HEC-RAS study MIDFKRIV.prj: MIDFKRIV

--- MIDFKRIV.g01 (geometry) --- (continued)

Type RM Length L Ch R = 1 ,101609  ,403.8,403.8,403.8
XS GIS Cut Line= 2
2243959.13670186648954.9663820432244393.10864511 649417.55576079
#Sta/Elev= 30
       0 2190.78    10.8  2188.9    19.5 2183.97    30.5 2180.27    52.4  2174.9
    83.4 2169.43   107.2 2161.65   121.2 2160.01   132.5 2160.83   146.6 2166.15
   152.3 2167.42   177.8 2167.79     195 2169.16   228.7  2169.5   271.1 2168.98
   310.2  2166.7   319.2 2165.05   330.6 2164.36  339.722161.657   348.6 2160.09
   398.5 2160.43  416.372161.674   425.4 2163.76   457.9 2192.52   463.7  2196.3
   491.9 2200.42   518.6 2208.78   548.5 2210.02   562.6 2215.14   634.3 2229.86
#Mann= 5 ,-1,0
       0      .1       0  339.72    .045       0  416.37      .1       0
     510     .06       0     560      .1       0
#XS Ineff= 2 , 0
          195.48 2174.42
Permanent Ineff=
       F       F
Bank Sta=339.72,416.37
XS Rating Curve= 0 ,0
Exp/Cntr(USF)=0,0
Exp/Cntr=0.3,0.1

Type RM Length L Ch R = 1 ,101205  ,344.8,344.8,344.8
XS GIS Cut Line= 2
2243661.70560759649109.4647008362244035.28466721649658.397196596
#Sta/Elev= 30
       0 2209.65    67.4 2185.93    76.4 2181.68    86.7 2180.91    96.4 2177.06
   130.3 2168.92   145.5 2166.04   177.2 2162.96   189.2 2159.16   202.9 2158.01
   222.2 2158.44   236.7 2162.07   254.9 2164.46   304.5 2167.17   321.1 2165.48
   338.5 2160.87   361.5 2163.05   401.2 2158.35   415.8  2157.1   459.3    2157
   475.82158.353   483.5 2160.84   494.9 2172.53   507.7 2181.91   528.4  2189.9
   557.2 2191.02   571.6 2196.61   623.5 2211.91   632.1 2212.96     664 2223.67
#Mann= 5 ,-1,0
       0      .1       0   401.2    .045       0   475.8      .1       0
     500     .06       0     620      .1       0
#XS Ineff= 2 , 0
          303.02 2186.69
Permanent Ineff=
       F       F
Bank Sta=401.2,475.8
XS Rating Curve= 0 ,0
Exp/Cntr(USF)=0,0
Exp/Cntr=0.3,0.1

Type RM Length L Ch R = 1 ,100860  ,220.6,220.6,220.6
XS GIS Cut Line= 2
2243394.86909085649341.5014639112243740.66714955649831.831661434
#Sta/Elev= 30
       0 2203.49    17.9 2201.28    57.8 2191.59    71.7 2185.44    82.8 2182.23
   112.2 2168.83   132.7 2157.47   175.8 2156.28   185.6 2157.15   195.4  2160.6
   210.1 2161.24   229.7 2159.91   253.3 2160.94   268.8  2158.8     305 2160.49
   328.5 2159.12   342.2 2159.94   350.9 2157.77   386.3 2156.42  426.062157.831
   435.2 2164.17   454.8 2169.26   468.6 2178.28   494.4 2179.32   503.8 2184.58
   531.7 2194.24   542.9 2200.95   560.4 2203.65   582.1 2213.98     600 2220.01
#Mann= 5 ,-1,0
       0      .1       0   350.9    .045       0  426.06      .1       0
     470     .06       0     590      .1       0
Bank Sta=350.9,426.06
XS Rating Curve= 0 ,0
Exp/Cntr(USF)=0,0
Exp/Cntr=0.3,0.1

Type RM Length L Ch R = 1 ,100640  ,49.4,49.4,49.4
XS GIS Cut Line= 2
2243271.50701584 649383.062854062243540.62469312650036.567834961
#Sta/Elev= 30
       0 2204.88    17.5 2197.67    28.2  2196.4    45.5 2190.51    54.2 2188.65
    75.8 2184.76    84.5 2184.61   124.7 2179.35   152.3 2171.77   179.7  2157.4
   195.2 2155.69   222.9 2157.67   265.6 2158.32   296.4  2156.5   339.7 2155.91
   391.3 2156.82   431.1 2156.83   469.5 2158.88   477.1  2160.9   499.8 2172.88
   525.7 2173.16     543    2181     556 2184.04     582 2192.96   599.3 2200.77
   612.2  2201.9   633.9 2212.66   645.6 2214.68   663.5 2223.41   706.7 2240.29
#Mann= 5 ,-1,0
       0      .1       0   391.3    .045       0   431.1      .1       0
     470     .06       0     580      .1       0
Bank Sta=391.3,431.1
XS Rating Curve= 0 ,0
Exp/Cntr(USF)=0,0
Exp/Cntr=0.3,0.1

Type RM Length L Ch R = 1 ,100590  ,181.7,181.7,181.7
XS GIS Cut Line= 2
2243226.46653422649403.2525502632243495.58421149650056.757531164
#Sta/Elev= 30
       0 2209.02    24.2 2196.43    39.6 2195.48    71.3 2184.96   149.2  2173.7
   159.1 2169.96   175.1 2160.04   186.6 2156.37   201.9 2155.29   235.7 2158.65
   244.3 2158.28   257.3 2154.94   303.1 2157.53   315.3 2157.37   330.1 2154.84
   375.5 2154.67   403.7 2154.04   434.7 2154.68   460.6 2157.46   477.7 2164.57
   495.2 2167.11   505.3 2171.95   534.2  2172.4   568.8 2184.49   603.3 2199.78
   620.7 2202.64   633.7 2211.09   642.3 2213.46   676.9 2228.32   706.7 2237.91
#Mann= 5 ,-1,0
       0      .1       0   375.5    .045       0   434.7      .1       0
     450     .06       0     600      .1       0
Bank Sta=375.5,434.7
XS Rating Curve= 0 ,0
Exp/Cntr(USF)=0,0
Exp/Cntr=0.3,0.1

Type RM Length L Ch R = 1 ,100409  ,387.4,387.4,387.4
XS GIS Cut Line= 4
2243037.48765509649490.1623195812243211.15896921649757.896357695
2243206.15682184649891.7037997792243380.68335711650096.850079516
#Sta/Elev= 30
       0 2215.85    47.5 2194.89      56 2193.41    75.1 2195.58    85.8 2194.37
   108.5 2183.17   137.1 2177.58   156.2 2170.85     169 2164.17   199.1 2161.86
   212.3 2153.51   261.1 2157.02   294.4 2154.32   319.1 2156.09     329 2153.71
   369.3 2152.29  412.312153.729   421.6  2156.8     455 2161.82   474.7  2157.5
   512.7 2157.67   528.5 2161.48   542.6 2167.89   571.8 2167.83   591.5 2179.65
   651.3 2199.96   665.5 2206.46   682.5 2208.05   699.5  2216.9   722.4 2225.38
#Mann= 5 ,-1,0
       0      .1       0     329    .045       0  412.31      .1       0
  483.03     .06       0  613.03      .1       0
#XS Ineff= 2 , 0
                           456.3         2166.38
Permanent Ineff=
       F       F
Bank Sta=329,412.31
XS Rating Curve= 0 ,0
Exp/Cntr(USF)=0,0
Exp/Cntr=0.3,0.1

Type RM Length L Ch R = 1 ,100021  ,357.5,357.5,357.5
XS GIS Cut Line= 2
2242662.95342781649742.2618834492243169.95358014650235.919926511
#Sta/Elev= 30
       0 2216.52    12.9 2215.75    22.7 2210.29    53.8 2199.85    70.8 2192.29
   101.7 2191.16   107.6 2187.64   146.9 2175.86   169.8 2167.01   216.3 2156.21
  227.572149.707   233.5 2147.68   267.9 2147.48  290.822149.704   299.9 2152.26
   314.3 2151.19   410.3 2156.57   469.7 2154.75   512.1 2156.82   526.5 2154.72
   537.5 2157.79   548.9 2157.78     560 2160.11   571.5 2160.89   594.8 2158.61
   599.1  2160.8   611.1 2171.76   670.5  2195.6   680.8  2197.4   707.6 2211.32
#Mann= 5 ,-1,0
       0      .1       0  227.57    .045       0  290.82      .1       0
     560     .06       0     700      .1       0
#XS Ineff= 2 , 0
                          410.18         2161.81
Permanent Ineff=
       F       F
Bank Sta=227.57,290.82
XS Rating Curve= 0 ,0
Exp/Cntr(USF)=0,0
Exp/Cntr=0.3,0.1

Type RM Length L Ch R = 1 ,99664   ,455.4,455.4,455.4
XS GIS Cut Line= 3
2242368.77318287649979.9820091172242818.51834618650366.912963399
2243061.91867063650448.694442102
#Sta/Elev= 30
       0 2209.59    50.9 2191.52    69.3 2187.44    82.7 2182.09   105.4 2181.83
   236.7 2166.46   241.9 2164.14  259.012148.012   264.2 2145.93   277.8 2145.57
   321.1 2145.72  329.722148.009   339.2 2151.59   351.4 2150.27     376 2151.61
   414.5 2150.62   458.3 2153.16   533.7 2153.54   576.2 2156.57   641.4 2154.19
   666.8 2154.65   700.5 2151.79   721.6 2153.36   751.2 2151.22   772.3 2148.03
     783 2149.99   789.1 2153.15   814.3  2174.1   831.3 2184.25   850.1 2187.66
#Mann= 5 ,-1,0
       0      .1       0  259.01    .045       0  329.72      .1       0
  643.28     .06       0  753.28      .1       0
#XS Ineff= 2 , 0
                          575.47         2161.81
Permanent Ineff=
       F       F
Bank Sta=259.01,329.72
XS Rating Curve= 0 ,0
Exp/Cntr(USF)=0,0
Exp/Cntr=0.3,0.1

Type RM Length L Ch R = 1 ,99208   ,547.6,547.6,547.6
XS GIS Cut Line= 3
2242142.99295801650516.5303802652242903.23015108 650618.93058298
2243045.19858749650594.447493206
#Sta/Elev= 30
       0  2191.7    57.7 2180.75    73.8 2179.72    81.9 2177.97      94 2178.09
   110.2  2180.9   154.6 2165.13   162.6 2156.74   174.7 2146.82  178.242145.056
   243.4 2143.22  266.272145.053   275.6 2148.51   372.5 2150.91   400.8 2153.58
   420.9 2152.31   445.2    2154   550.1 2153.46   558.2 2154.57   567.2 2152.98
   590.5 2153.16   691.4 2149.51   719.6 2150.12   800.6  2148.5   812.7 2150.34
   845.2 2146.66   853.3 2149.95   873.6 2163.04     898  2176.7   911.2 2185.84
#Mann= 5 ,-1,0
       0      .1       0  178.24    .045       0  266.27      .1       0
   827.1     .06       0   867.1      .1       0
#XS Ineff= 2 , 0
                          557.38         2158.69
Permanent Ineff=
       F       F
Bank Sta=178.24,266.27
XS Rating Curve= 0 ,0
Exp/Cntr(USF)=0,0
Exp/Cntr=0.3,0.1

Type RM Length L Ch R = 1 ,98661   ,534.2,534.2,534.2
XS GIS Cut Line= 3
2242311.78787424 651135.087918572242638.50576077650862.477022071
2243065.29638642650655.647168446
#Sta/Elev= 30
       0 2192.06    52.6  2173.6    73.4 2173.51    78.6  2169.2    89.1 2152.39
   98.882141.913   104.7 2140.04   149.3 2140.53   182.8 2139.43  189.912141.916
   197.6  2145.7   208.9 2147.59   271.5 2145.03   292.2 2146.13     314 2149.51
   333.9 2150.63   352.6 2149.91     368 2151.69   425.5  2149.7   458.5 2150.48
   492.7 2148.93   643.3  2148.8   725.2 2147.29     743    2149   778.5 2147.11
     790 2149.09   818.5 2147.48   849.9 2152.46   880.8  2169.8   899.8 2182.27
#Mann= 5 ,-1,0
       0      .1       0   98.88    .045       0  189.91      .1       0
  785.51     .06       0  895.51      .1       0
#XS Ineff= 2 , 0
                          211.42         2152.69
Permanent Ineff=
       F       F
Bank Sta=98.88,189.91
XS Rating Curve= 0 ,0
Exp/Cntr(USF)=0,0
Exp/Cntr=0.3,0.1

Type RM Length L Ch R = 1 ,98127   ,466.6,466.6,466.6
XS GIS Cut Line= 3
2242718.63267196651535.9788756622243087.47832674 650962.01339283
2243280.95035995650824.077055869
#Sta/Elev= 30
       0  2173.1    69.7 2151.53   107.3 2143.97   130.5 2143.72  140.392137.752
   193.5 2136.26  210.732137.754   236.3 2141.68   295.5 2138.26   315.8 2142.94
   350.4 2143.01   362.1 2140.91     379 2142.39   431.3 2141.53   483.8 2138.57
   528.2 2143.69     640 2144.44   651.5 2142.67   678.5 2142.61     692 2145.98
   760.8 2144.54   776.5 2147.15   786.6 2152.54   800.9 2163.73   815.3 2167.62
   841.1 2187.22   862.9 2199.33   874.7 2201.47   884.5 2209.08   919.9 2229.33
#Mann= 5 ,-1,0
       0      .1       0  140.39    .045       0  210.73      .1       0
     640     .06       0  772.26      .1       0
#XS Ineff= 2 , 0
                          345.96            2150
Permanent Ineff=
       F       F
Bank Sta=140.39,210.73
XS Rating Curve= 0 ,0
Exp/Cntr(USF)=0,0
Exp/Cntr=0.3,0.1

Type RM Length L Ch R = 1 ,97660   ,361.6,361.6,361.6
XS GIS Cut Line= 4
2242839.21095378651777.3208538192243184.89690238651679.945939369
2243237.84178044651582.5273637322243577.93451701651256.808553146
#Sta/Elev= 30
       0 2183.68      43 2164.27    96.6 2143.46     109 2140.98   125.7 2139.34
   183.9 2140.37   204.6 2145.83   225.4 2140.46   271.1 2138.36   371.4 2140.12
   384.2 2132.56   391.1 2131.32   446.2 2132.53   466.5 2136.78   498.1 2137.29
   577.3 2134.37   593.4 2131.44   633.9 2136.47   697.5 2135.61   720.6 2133.28
   732.2 2136.99   749.9 2135.41     764 2144.58   794.5 2143.66   805.6 2148.22
   833.3 2152.18   859.4 2161.71     872 2163.44   911.5 2180.27   940.9 2196.32
#Mann= 5 ,-1,0
       0      .1       0   384.2    .045       0   446.2      .1       0
  750.01     .06       0  890.01      .1       0
#XS Ineff= 2 , 0
                          736.57         2139.76
Permanent Ineff=
       F       F
Bank Sta=384.2,446.2
XS Rating Curve= 0 ,0
Exp/Cntr(USF)=0,0
Exp/Cntr=0.3,0.1

Type RM Length L Ch R = 1 ,97298   ,472.1,472.1,472.1
XS GIS Cut Line= 4
2243177.44200793652424.249348486 2243534.3330976651807.013646721
2243568.21781956651694.7705052262243786.25708078651531.827743571
#Sta/Elev= 30
       0 2209.28    26.6  2193.2    63.6 2175.32    77.5 2174.08   119.1 2161.91
   142.2  2152.5   160.6 2142.15   171.1 2139.38   243.8 2137.05   301.1  2138.1
   350.1 2135.64   391.7 2136.99   419.4 2134.43   575.1 2131.72   604.8 2136.93
   618.1 2135.57   627.8 2131.25   642.5 2129.12   687.4 2132.67   723.3 2131.73
  733.832129.553   805.8 2129.57   880.1 2132.07   900.1 2127.61   925.6 2140.82
     950 2145.62   966.5 2160.12  1009.9 2161.91  1029.9 2172.64  1102.4 2191.47
#Mann= 5 ,-1,0
       0      .1       0  733.83    .045       0   805.8      .1       0
  850.23     .06       0 1010.23      .1       0
#XS Ineff= 2 , 0
          685.13 2137.96
Permanent Ineff=
       F       F
Bank Sta=733.83,805.8
XS Rating Curve= 0 ,0
Exp/Cntr(USF)=0,0
Exp/Cntr=0.3,0.1

Type RM Length L Ch R = 1 ,96826   ,387.8,387.8,387.8
XS GIS Cut Line= 3
2243327.26500053652456.7151474312243499.13103677652251.951732013
2244121.38141104651959.890347345
#Sta/Elev= 30
       0 2183.38    15.1 2178.68    51.4 2162.51    62.8 2161.97    99.7  2143.7
   124.7 2135.48   139.4 2134.63   156.5 2135.74   190.5 2134.06   330.3 2132.09
   396.2 2132.29   409.9 2129.61   519.8  2128.9   529.2 2127.58   537.8 2123.78
   542.4 2123.28   560.1 2125.17   573.4 2123.84  661.322125.155   666.2 2128.32
     675  2136.7   679.4 2139.35   692.7 2139.84   703.2 2144.56   718.3 2148.45
   745.7 2146.98     759 2149.82   834.1 2150.28   922.5 2159.57   954.7 2166.14
#Mann= 6 ,-1,0
       0      .1       0  437.33     .05       0  447.33      .1       0
   560.1    .045       0  661.32     .06       0  767.33      .1       0
#XS Ineff= 2 , 0
          557.38 2135.92
Permanent Ineff=
       F       F
Bank Sta=560.1,661.32
XS Rating Curve= 0 ,0
Exp/Cntr(USF)=0,0
Exp/Cntr=0.3,0.1

Type RM Length L Ch R = 1 ,96439   ,515.4,515.4,515.4
XS GIS Cut Line= 2
 2243619.0922337652658.6755345922244214.64275968652272.602715273
#Sta/Elev= 30
       0  2165.3    15.6 2156.22    32.2 2141.46    42.4 2130.85    46.9  2128.3
      51  2127.5    77.6 2125.87   163.4 2125.03   182.4 2127.69   225.3  2129.5
   282.5 2129.47   333.7 2127.31     354 2128.86   360.5 2127.74   373.22122.667
   377.8 2120.94   399.8 2120.46  434.282122.677     482 2122.42   496.4 2126.52
   520.9 2128.54   539.6 2127.94     560 2132.36   571.6 2133.24   587.6 2137.34
   613.1 2136.86   630.5 2138.91   644.8 2138.64   676.2 2142.67   709.7 2145.28
#Mann= 6 ,-1,0
       0      .1       0     280     .05       0   373.2    .045       0
  434.28      .1       0     530     .06       0  709.74      .1       0
#XS Ineff= 2 , 0
          225.66 2134.82
Permanent Ineff=
       F       F
Bank Sta=373.2,434.28
XS Rating Curve= 0 ,0
Exp/Cntr(USF)=0,0
Exp/Cntr=0.3,0.1

Type RM Length L Ch R = 1 ,95923   ,633.2,633.2,633.2
XS GIS Cut Line= 2
2244013.91664064653054.4357455482244523.47958206652625.129403068
#Sta/Elev= 30
       0 2173.89    13.8 2157.02      33 2143.94    45.4 2130.45    51.6 2127.66
    62.1 2125.75    70.9 2120.81    88.9 2119.76   101.3 2120.21   112.8 2122.51
   215.4 2124.67   227.9 2123.75   238.3 2118.47   243.6 2117.13   255.1 2117.02
   294.9 2117.22   303.4 2118.42     322 2122.25     346 2120.52   391.4 2123.12
   437.1  2122.7   453.9 2124.14     511 2125.52     526 2127.66   536.5  2131.1
   567.8 2128.82   575.9 2131.58   588.8 2131.85   651.5  2143.4   666.3 2147.23
#Mann= 5 ,-1,0
       0      .1       0   238.3    .045       0   303.4      .1       0
     430     .06       0     600      .1       0
#XS Ineff= 2 , 0
          212.49 2129.26  392.54         2127.06
Permanent Ineff=
       F       F
Bank Sta=238.3,303.4
XS Rating Curve= 0 ,0
Exp/Cntr(USF)=0,0
Exp/Cntr=0.3,0.1

Type RM Length L Ch R = 1 ,95290   ,308.3,308.3,308.3
XS GIS Cut Line= 2
2244440.54887624653496.9599017232244987.80019917653087.833223232
#Sta/Elev= 30
       0 2156.13    14.5 2150.99    45.3 2136.78    59.8 2133.31    88.2 2119.21
   116.7 2119.11     131 2115.24   139.6 2117.44   146.6 2115.79   154.4 2114.62
   219.3 2114.76   224.92115.845   233.9 2117.79   320.3 2117.19   333.7 2114.12
   353.9 2113.56   365.4 2114.17   374.1 2117.17   404.1 2117.25   462.5 2125.44
   523.9 2130.95   533.9  2135.6   545.4 2137.76   583.9 2139.94   605.4 2143.22
   633.8 2152.83   642.6 2150.59   665.4 2151.91   676.9 2157.57   683.3 2159.21
#Mann= 4 ,-1,0
       0      .1       0   146.6    .045       0   224.9      .1       0
     560     .06       0
Bank Sta=146.6,224.9
XS Rating Curve= 0 ,0
Exp/Cntr(USF)=0,0
Exp/Cntr=0.3,0.1

Type RM Length L Ch R = 1 ,94982   ,278.7,278.7,278.7
XS GIS Cut Line= 3
2244519.59859301653684.2858109952245048.17517795653583.966891103
2245171.41653157653464.449964023
#Sta/Elev= 30
       0 2140.75      25 2127.86    49.4 2120.37    78.4 2118.87   204.2 2118.65
   208.5 2117.89   216.4 2112.96   224.5 2111.04   265.2  2110.8  276.182112.985
   285.6 2116.93   330.4 2117.41   403.5 2115.75   415.9  2116.7   424.1 2115.44
   436.2 2117.05     448    2116   467.2 2111.52   475.4 2113.42   485.1 2118.95
   493.2 2121.26   533.6 2123.62   553.5 2126.32   582.2 2125.07   636.2 2126.32
     655 2128.92   666.2 2134.38   688.5 2135.18   699.6 2133.89   709.7 2137.61
#Mann= 6 ,-1,0
       0      .1       0     120     .06       0     160     .05       0
   216.4    .045       0  276.18      .1       0  648.01     .07       0
Bank Sta=216.4,276.18
XS Rating Curve= 0 ,0
Exp/Cntr(USF)=0,0
Exp/Cntr=0.3,0.1

Type RM Length L Ch R = 1 ,94703   ,126.1,126.1,126.1
XS GIS Cut Line= 3
2244553.69944452653887.131611048 2245084.9900218653896.898303783
2245235.25140316654020.131146127
#Sta/Elev= 30
       0 2139.79    26.5 2122.54    34.5  2119.2    50.5 2114.95   194.5 2118.37
   210.5 2116.95   226.5 2117.02   238.5 2113.79   253.1 2112.09   266.5 2110.69
   314.5 2110.75  321.582112.106   334.4 2114.38   350.5 2115.59   374.5 2114.39
   399.8 2116.02   414.5 2115.63   430.5    2118   450.6 2119.18   483.7 2118.99
   498.6 2120.98   518.6 2126.36   562.3 2127.07   619.1  2132.4   633.8 2132.29
   680.3 2135.18   690.7 2136.44   695.9 2137.94   706.2 2144.04   725.7 2146.18
#Mann= 8 ,-1,0
       0      .1       0      90     .06       0     180     .05       0
   253.1    .045       0  321.58      .1       0  591.38     .06       0
  621.38      .1       0  721.38     .06       0
#XS Ineff= 2 , 0
          195.36 2120.85
Permanent Ineff=
       F       F
Bank Sta=253.1,321.58
XS Rating Curve= 0 ,0
Exp/Cntr(USF)=0,0
Exp/Cntr=0.3,0.1

Type RM Length L Ch R = 1 ,94577   ,46.8,46.8,46.8
XS GIS Cut Line= 2
2244540.15143233653913.0792965072245227.93419001654164.287137308
#Sta/Elev= 30
       0 2147.65     8.5 2140.82    40.6 2120.43    46.9 2117.81    56.2 2116.27
    80.9 2114.39   112.4 2116.19   200.2 2116.78   221.5 2114.77   242.8 2114.21
  258.482112.021   265.2 2110.74   306.6 2110.66   332.2  2110.7   346.3 2113.37
   373.4  2111.6  388.752112.022   483.6 2115.22   498.3 2116.45   536.6 2115.47
   545.1 2116.42   549.4 2117.35   562.1 2125.42   570.7 2129.73   583.4 2132.95
   643.1 2139.51   681.4 2146.68   698.4 2150.63   708.2 2154.13   732.2 2157.44
#Mann= 8 ,-1,0
       0      .1       0     110     .06       0     210      .1       0
  258.48    .045       0  388.75      .1       0     400     .06       0
     630      .1       0     690     .06       0
#XS Ineff= 2 , 0
          164.61 2119.23
Permanent Ineff=
       F       F
Bank Sta=258.48,388.75
XS Rating Curve= 0 ,0
Exp/Cntr(USF)=0,0
Exp/Cntr=0.3,0.1

Type RM Length L Ch R = 1 ,94530   ,191,191,191
XS GIS Cut Line= 2
2244517.36039839653954.6096250272245205.14315606654205.817465828
#Sta/Elev= 30
       0 2155.89    11.5  2146.4    44.7 2123.61    57.2 2117.48    66.9 2114.58
    83.9 2113.62     129 2115.29     195 2115.95   213.2 2116.98   219.4 2115.96
   228.7 2112.43  238.422109.917   245.7 2108.09   279.8  2107.8     338 2107.96
   359.8 2108.88  365.372109.917   378.5 2113.78   484.2 2112.94   520.5 2115.95
   535.3 2115.75   548.1 2114.53   586.4 2115.89   590.7 2116.87   594.9  2118.9
   620.5 2133.96   671.6 2143.07   709.9 2153.63   722.7 2158.03   732.2 2159.44
#Mann= 6 ,-1,0
       0      .1       0     130     .06       0  238.42    .045       0
  365.37     .06       0     560      .1       0     650     .06       0
#XS Ineff= 2 , 0
          211.19 2121.63
Permanent Ineff=
       F       F
Bank Sta=238.42,365.37
XS Rating Curve= 0 ,0
Exp/Cntr(USF)=0,0
Exp/Cntr=0.3,0.1

Type RM Length L Ch R = 1 ,94339   ,470.2,470.2,470.2
XS GIS Cut Line= 2
2244406.94255763654116.9970793692245128.62830115654381.745152274
#Sta/Elev= 30
       0 2160.98    23.8 2147.22    44.7 2140.59    57.2 2131.21      79 2118.55
    90.8 2114.23   103.6 2112.65   116.4 2109.29   153.8 2108.54   167.5 2110.88
   201.6 2110.73   222.9 2109.25     244 2111.15   269.7 2110.44   312.8 2111.69
  330.352107.598   354.9 2106.28   380.5 2106.42     3872107.531   401.8 2111.39
   521.1 2112.24   550.9  2113.8   593.4 2111.32   606.3 2112.69   648.9 2110.41
   670.2 2110.89   674.5 2112.46     683 2118.36     718 2147.99   768.7 2161.76
#Mann= 4 ,-1,0
       0      .1       0  330.35    .045       0     387      .1       0
  768.71     .06       0
Bank Sta=330.35,387
XS Rating Curve= 0 ,0
Exp/Cntr(USF)=0,0
Exp/Cntr=0.3,0.1

Type RM Length L Ch R = 1 ,93869   ,367.6,367.6,367.6
XS GIS Cut Line= 2
 2244288.2199106654575.9348529722245020.32130312 654838.89186833
#Sta/Elev= 30
       0 2140.93    12.7  2138.1      76 2130.77      85 2128.57   123.2 2126.29
   178.5 2119.47   191.2 2113.05   199.7 2111.65  213.842105.496     221 2104.34
     255 2104.22     356 2105.49   382.4 2108.22     425 2107.89   501.5 2103.12
   518.5 2105.69   535.7 2104.54   554.4 2105.93   607.6 2103.92   624.7 2106.59
     642 2104.57   663.9 2106.02   671.5 2109.93   688.5 2124.65   692.7 2131.32
   704.5 2153.99     714 2162.81   757.7  2192.2   763.9 2193.95   777.9 2194.49
#Mann= 4 ,-1,0
       0      .1       0  213.84    .045       0     356      .1       0
     770     .06       0
Bank Sta=213.84,356
XS Rating Curve= 0 ,0
Exp/Cntr(USF)=0,0
Exp/Cntr=0.3,0.1

Type RM Length L Ch R = 1 ,93501   ,486.8,486.8,486.8
XS GIS Cut Line= 2
2244283.50193785655019.4922914882244907.38512199655035.360680776
#Sta/Elev= 30
       0 2133.27    96.7 2118.13   196.7 2109.55   204.7 2106.87   212.7 2106.35
   223.92101.952   232.7 2100.42   267.6 2100.29   284.8 2100.55   292.8 2102.01
   312.8 2104.23   364.8 2103.99     389 2106.79   432.8 2106.47   456.8 2104.42
   464.8 2101.51   484.8 2099.59   508.8 2103.56   521.3 2103.71   529.1 2106.84
   540.8 2117.72   556.9  2130.4   569.7  2143.7   572.9 2147.69   580.9 2167.28
   584.9 2175.54   588.9 2179.61   604.9 2190.42   616.9 2193.27   624.1 2193.48
#Mann= 4 ,-1,0
       0      .1       0   223.9    .045       0   292.8      .1       0
     550     .06       0
Bank Sta=223.9,292.8
XS Rating Curve= 0 ,0
Exp/Cntr(USF)=0,0
Exp/Cntr=0.3,0.1

Type RM Length L Ch R = 1 ,93014   ,483.6,483.6,483.6
XS GIS Cut Line= 2
2244226.80588238655490.6989660672244795.64376408655522.987779993
#Sta/Elev= 30
       0  2138.4    89.5 2120.22   125.6 2114.25   133.6 2111.31   149.6  2101.2
   157.6 2099.51   161.6 2099.47   170.5 2101.45   181.7 2101.56   193.2 2103.92
   209.7 2101.78   241.8 2102.56   250.1 2103.73   272.8 2101.07   297.8 2101.31
   305.9 2100.46   312.22098.474   322.1 2096.64   337.9 2095.93     379 2096.16
  390.562098.472     406 2103.15   462.1 2105.91   466.2 2107.06   510.2 2134.38
   514.2 2135.87   526.2 2137.08   534.2 2142.67   553.4 2151.66   569.8 2161.97
#Mann= 3 ,-1,0
       0      .1       0   312.2    .045       0  390.56      .1       0
Bank Sta=312.2,390.56
XS Rating Curve= 0 ,0
Exp/Cntr(USF)=0,0
Exp/Cntr=0.3,0.1

Type RM Length L Ch R = 1 ,92531   ,412.7,412.7,412.7
XS GIS Cut Line= 2
2244215.88339426655935.510846028 2244800.0040425655900.551293745
#Sta/Elev= 30
       0 2149.22    31.9 2137.32    40.4 2131.95    48.4 2131.97    52.4 2129.36
    68.4 2114.49   91.422096.193   100.5 2093.77   124.5 2093.56   148.6  2093.7
  162.262096.195   172.6 2099.57   176.6 2099.89   188.6 2100.18   204.7  2098.9
   212.7 2102.98   216.7 2102.89   228.7 2099.12   236.7  2098.1   284.8 2099.97
   304.8 2099.44   364.9 2103.98     397 2102.11   440.8  2101.9   481.2 2118.49
   516.7 2128.22   541.3 2137.52   553.3 2138.86   565.3  2143.9   585.2 2148.76
#Mann= 3 ,-1,0
       0      .1       0   91.42    .045       0  162.26      .1       0
#XS Ineff= 1 ,-1
  365.03585.1659 2110.58
Permanent Ineff=
       F
Bank Sta=91.42,162.26
XS Rating Curve= 0 ,0
Exp/Cntr(USF)=0,0
Exp/Cntr=0.3,0.1

Type RM Length L Ch R = 1 ,92118   ,423.7,423.7,423.7
XS GIS Cut Line= 3
2244237.43152471656349.7894204632244719.63119657656307.933543236
2244864.23517145656212.233149265
#Sta/Elev= 30
       0  2158.9     6.8 2152.84    34.9 2136.51      63 2115.56      71 2108.27
      79 2103.95   94.542093.862    99.1 2092.39   103.1 2092.12   150.9 2091.95
   171.4 2092.05  192.392093.863   223.6 2096.94   247.7 2098.13   259.7 2097.64
   271.8 2099.11   283.8 2099.47   360.1 2097.29   376.2 2097.88   384.2 2097.32
   400.2 2098.11   412.3 2096.76   420.3 2096.82   428.3 2098.56   436.4 2102.28
   440.4 2103.27   497.9 2107.86   538.3 2112.02   638.2 2126.27   657.4 2130.26
#Mann= 3 ,-1,0
       0      .1       0   94.54    .045       0  192.39      .1       0
#XS Ineff= 2 , 0
                          287.28         2104.51
Permanent Ineff=
       F       F
Bank Sta=94.54,192.39
XS Rating Curve= 0 ,0
Exp/Cntr(USF)=0,0
Exp/Cntr=0.3,0.1

Type RM Length L Ch R = 1 ,91694   ,506.3,506.3,506.3
XS GIS Cut Line= 3
2244234.42506452656790.9439748372245046.27733075656657.838587499
2245162.24376483656577.664952656
#Sta/Elev= 30
       0 2196.72    13.9 2195.23    38.3 2185.91    50.4 2173.93    74.7 2138.63
   127.4 2095.06  140.362091.628   155.8 2089.72   200.4 2089.58   236.9 2089.72
   244.82091.627   253.1 2094.23   292.1 2093.34   317.9 2097.82   366.6  2096.9
   431.4 2092.03   476.7 2092.87   581.8 2097.17   675.2 2104.62   694.9 2104.48
   739.5 2107.73   771.9  2111.6   788.1 2117.79   796.2 2119.35   816.5 2120.67
   844.4 2119.56     859 2123.47   902.2 2129.04   916.5 2138.67   963.7 2157.76
#Mann= 6 ,-1,0
       0      .1       0  140.36    .045       0   244.8      .1       0
     530     .05       0     810     .06       0  922.69      .1       0
#XS Ineff= 2 , 0
                          333.33         2127.49
Permanent Ineff=
       F       F
Bank Sta=140.36,244.8
XS Rating Curve= 0 ,0
Exp/Cntr(USF)=0,0
Exp/Cntr=0.3,0.1

Type RM Length L Ch R = 1 ,91188   ,452.5,452.5,452.5
XS GIS Cut Line= 4
2244335.24605185657228.0511803012244434.53841053 657270.02291286
2245064.09536661 657155.090171562245183.63120495657202.130048163
#Sta/Elev= 30
       0 2160.79    27.1 2146.37    66.1 2114.15    74.8 2108.62    85.1 2104.48
    99.2 2097.14   113.5 2091.52  139.162088.035   150.1 2086.75   211.1 2086.82
   216.5 2088.03   223.3 2089.38   255.8 2090.54   340.3 2090.14   369.7 2088.88
   406.3 2089.06   426.6 2085.88   442.9 2089.15   467.3 2091.21   577.1 2094.82
   598.2 2096.69   642.1 2103.12   670.4 2108.78   708.2 2110.06   718.5 2111.93
   731.6 2116.01   769.3 2117.88   812.3 2122.46   842.4 2131.56   876.2 2139.14
#Mann= 6 ,-1,0
       0      .1       0  139.16    .045       0   216.5      .1       0
   617.8     .05       0   717.8     .07       0  817.76      .1       0
Bank Sta=139.16,216.5
XS Rating Curve= 0 ,0
Exp/Cntr(USF)=0,0
Exp/Cntr=0.3,0.1

Type RM Length L Ch R = 1 ,90736   ,459.5,459.5,459.5
XS GIS Cut Line= 3
2244187.25766014657608.6725262192244327.51884412 657704.24115754
2245028.40707704657689.643116404
#Sta/Elev= 30
       0 2142.81    86.1 2107.23   107.5 2100.34   135.9  2093.6   283.1 2093.02
   326.2 2090.41   382.4 2089.96   386.4 2089.14  393.672084.892     441 2083.53
   472.22084.823   486.4 2086.34   542.5 2086.28   582.5 2085.06   610.5 2081.62
   638.5 2082.86   666.5  2099.8   670.5 2101.34   682.5 2098.08   690.3 2099.19
   706.5 2109.89   710.5 2111.27   782.5 2113.11   790.5 2116.11   798.5 2116.79
   806.5 2119.67   827.9 2123.51   850.5 2130.81   859.2 2131.52   870.8 2135.04
#Mann= 6 ,-1,0
       0     .05       0  379.72      .1       0  393.67    .045       0
   472.2      .1       0  679.72     .06       0  859.72      .1       0
Bank Sta=393.67,472.2
XS Rating Curve= 0 ,0
Exp/Cntr(USF)=0,0
Exp/Cntr=0.3,0.1

Type RM Length L Ch R = 1 ,90276   ,413.7,413.7,413.7
XS GIS Cut Line= 3
2244039.32200397657780.1094176812244405.07301921658052.968880385
2244879.43894353658206.205864934
#Sta/Elev= 30
       0 2142.99      26 2130.63      46 2123.95    75.4 2112.13    95.7    2102
     110 2099.53   125.8 2093.32   130.8 2092.41   207.2 2088.91     468 2090.31
   528.8 2088.76   560.6 2089.43   602.5 2084.73   662.3 2083.63   682.4 2082.53
  689.582081.021   703.4 2078.89   749.6 2079.28  755.732081.021   773.5 2089.31
   800.1 2105.57   812.7 2107.84   825.3 2104.88   833.7 2105.21   846.3 2114.09
   859.3 2117.94     891 2119.86   896.7 2123.82   906.9 2127.48   954.8 2139.72
#Mann= 7 ,-1,0
       0      .1       0      20     .05       0  596.32      .1       0
  689.58    .045       0  755.73      .1       0  806.32     .06       0
  906.32      .1       0
Bank Sta=689.58,755.73
XS Rating Curve= 0 ,0
Exp/Cntr(USF)=0,0
Exp/Cntr=0.3,0.1

Type RM Length L Ch R = 1 ,89862   ,402.9,402.9,402.9
XS GIS Cut Line= 2
2243906.69058463657930.5564280852244567.32599917658627.977891695
#Sta/Elev= 30
       0 2152.72    17.1 2142.33    28.4 2138.27    53.2 2123.96    91.8 2106.03
    99.1 2101.37   112.7 2098.68   119.3 2094.35   146.9 2084.44   432.6 2088.08
   577.3    2087   619.7  2088.7   676.9 2085.87   690.5 2083.27  699.052078.718
     706 2076.14   730.1 2075.92     764  2076.4  772.252078.717   783.8 2081.83
   792.3 2081.65   806.5  2078.8   824.6  2081.1   830.1 2084.26   857.4 2104.89
   874.6  2109.9   890.7 2122.88   923.7 2125.38   940.3 2136.86   960.6 2142.66
#Mann= 7 ,-1,0
       0      .1       0     220     .05       0     630      .1       0
  699.05    .045       0  772.25      .1       0     890     .06       0
     920      .1       0
#XS Ineff= 2 , 0
          306.95 2098.69
Permanent Ineff=
       F       F
Bank Sta=699.05,772.25
XS Rating Curve= 0 ,0
Exp/Cntr(USF)=0,0
Exp/Cntr=0.3,0.1

Type RM Length L Ch R = 1 ,89460   ,425.4,425.4,425.4
XS GIS Cut Line= 2
2243656.70025804658119.3103401062244213.49457448658857.656914538
#Sta/Elev= 30
       0 2152.31    32.3 2128.24    85.5 2091.37    98.1 2089.06   106.6 2086.17
   132.6  2083.9   238.3 2079.05   252.8 2081.03     298    2083   490.7 2083.83
   548.4 2085.03   553.4 2084.71   568.5 2079.15   573.5 2078.59   646.4 2080.27
  656.062076.922   663.5 2075.07     675 2074.52   718.8 2074.64  730.262076.926
   748.8  2090.8     755  2094.1   788.9  2098.8   798.9 2103.02   820.7 2103.15
     834 2104.98   846.4 2107.93     859 2108.61   902.6 2115.64   924.8 2120.41
#Mann= 6 ,-1,0
       0      .1       0     210     .05       0     450      .1       0
  656.06    .045       0  730.26     .06       0     820      .1       0
#XS Ineff= 2 , 0
          345.96  2094.8
Permanent Ineff=
       F       F
Bank Sta=656.06,730.26
XS Rating Curve= 0 ,0
Exp/Cntr(USF)=0,0
Exp/Cntr=0.3,0.1

Type RM Length L Ch R = 1 ,89034   ,196.5,196.5,196.5
XS GIS Cut Line= 2
2243379.87124731658343.6633769792243822.39861121659011.458216974
#Sta/Elev= 30
       0 2124.84    16.2 2123.17    65.7 2111.75     111 2097.76     141 2094.05
   246.6 2087.57   266.8 2087.37   280.1 2089.81   294.5 2085.51   336.1 2083.04
   353.4  2077.1   379.4 2076.24   393.8 2072.85   400.1 2072.79   424.1    2078
   467.3 2077.08   480.4 2074.19   491.3 2072.42   520.1 2072.26   548.9 2072.42
  554.712074.136     568 2077.75   649.6 2077.36   702.4 2084.33   717.4 2089.36
   745.6 2089.05   755.2 2094.98   777.7 2102.55   789.8 2109.37   801.1 2111.69
#Mann= 6 ,-1,0
       0      .1       0      50     .05       0     400      .1       0
   480.4    .045       0  554.71      .1       0     670     .06       0
Bank Sta=480.4,554.71
XS Rating Curve= 0 ,0
Exp/Cntr(USF)=0,0
Exp/Cntr=0.3,0.1

Type RM Length L Ch R = 1 ,88838   ,45,45,45
XS GIS Cut Line= 4
2243240.07472421  658266.52145452243481.92370387658657.460000038
2243472.39362582658924.3021854762243674.98627414659182.978605639
#Sta/Elev= 30
       0 2104.56    15.4 2106.56    38.2 2104.33    77.6 2103.55   121.8 2098.41
   175.1 2098.75   251.9  2094.9   308.9 2089.77   337.1    2084   362.3 2085.51
   426.4 2082.68   463.4 2082.68   507.4 2078.09   575.5 2077.25   587.5 2075.71
   598.7  2072.3   615.3 2070.25   647.5 2070.31  658.862072.208   683.6 2076.55
   753.2 2073.94   819.3 2078.38   839.6  2078.6   858.2 2080.65   900.6 2080.73
   915.8 2084.85   941.2 2083.65   946.6  2085.5   983.6 2105.27  1055.3 2136.56
#Mann= 9 ,-1,0
       0      .1       0     140     .05       0     370     .06       0
     410     .05       0   479.7      .1       0   598.7    .045       0
  658.86      .1       0  786.71     .06       0  916.71      .1       0
Bank Sta=598.7,658.86
XS Rating Curve= 0 ,0
Exp/Cntr(USF)=0,0
Exp/Cntr=0.3,0.1

Type RM Length L Ch R = 1 ,88793   ,194.4,194.4,194.4
XS GIS Cut Line= 4
2243209.01046488658283.3020708592243441.32936649658657.086475905
2243431.79928844658923.9286613432243634.39193676659182.605081506
#Sta/Elev= 30
       0  2107.4    77.6 2103.43   152.9 2096.59   209.9 2096.66   218.9 2095.24
     233 2089.45   242.4 2088.26   270.7 2092.18   284.8 2092.34     346 2087.88
   448.2 2083.93   487.7 2078.03   520.2 2077.78   548.3 2075.02     576  2076.7
  591.312072.105   596.3 2070.54   612.3  2070.3   644.3 2070.38   652.3 2072.14
   660.3    2079   696.4 2075.87   762.4  2073.7   859.3 2079.98   910.6 2080.64
   922.1 2084.35   947.6 2082.95   967.6 2091.33  1013.5 2115.73  1035.7 2125.02
#Mann= 10 ,-1,0
       0      .1       0     120     .05       0     230     .06       0
     280     .05       0     350     .06       0  591.31    .045       0
   652.3     .06       0  747.11      .1       0  767.11     .06       0
  907.11      .1       0
Bank Sta=591.31,652.3
XS Rating Curve= 0 ,0
Exp/Cntr(USF)=0,0
Exp/Cntr=0.3,0.1

Type RM Length L Ch R = 1 ,88598   ,382.2,382.2,382.2
XS GIS Cut Line= 2
2243034.09665099658556.8019400162243500.68927238659320.161191931
#Sta/Elev= 30
       0 2114.56    36.7 2112.73     113 2113.49   126.9  2109.9   141.1 2103.15
   158.9 2091.95   173.9 2084.54   192.7 2077.94   298.6 2077.21   384.9 2078.14
  406.662071.868   414.9 2070.01   423.7 2069.47   450.5 2069.63  467.562071.867
   473.1 2074.56     476 2074.84   586.4  2072.6   595.8 2074.01   605.2 2073.21
   656.4 2078.08   717.3 2077.72   755.2 2081.09   781.6 2079.55   787.4 2081.97
   833.9 2111.18   844.3  2115.7     863 2126.88   870.7 2129.79   894.7 2142.89
#Mann= 7 ,-1,0
       0     .05       0      30      .1       0     260     .05       0
  406.66    .045       0  467.56      .1       0     490     .06       0
     810      .1       0
#XS Ineff= 2 ,-1
       0  383.85 2085.43  663.02894.6653 2087.07
Permanent Ineff=
       F       F
Bank Sta=406.66,467.56
XS Rating Curve= 0 ,0
Exp/Cntr(USF)=0,0
Exp/Cntr=0.3,0.1

Type RM Length L Ch R = 1 ,88216   ,469.5,469.5,469.5
XS GIS Cut Line= 3
2242683.21347544658631.0105679792242727.77928217658830.623249376
2243220.32463615659480.715860443
#Sta/Elev= 30
       0 2106.09    18.6 2100.56    30.9 2098.62   129.3 2076.78   198.9 2074.94
   298.1 2074.73   513.9 2077.17     575 2079.65   583.5 2078.51   594.2 2072.46
   599.2 2071.08   654.9 2071.52  672.782069.527   680.6 2067.55     712 2067.22
   734.7 2067.42   739.7 2069.52   760.5 2077.16   804.9 2077.02     815 2078.43
   826.2 2075.76   847.7 2074.07   874.2 2074.24   890.2 2077.13   905.3 2083.79
   935.4 2083.46   940.5 2086.96   971.8 2115.84  1005.7  2137.7  1020.1 2148.02
#Mann= 5 ,-1,0
       0      .1       0  672.78    .045       0   739.7      .1       0
  874.53     .06       0 1004.53      .1       0
#XS Ineff= 2 , 0
           394.8 2086.13   814.7         2083.99
Permanent Ineff=
       F       F
Bank Sta=672.78,739.7
XS Rating Curve= 0 ,0
Exp/Cntr(USF)=0,0
Exp/Cntr=0.3,0.1

Type RM Length L Ch R = 1 ,87747   ,407.5,407.5,407.5
XS GIS Cut Line= 4
2242180.22858777658962.3591357712242390.41451915659080.311294322
2242708.71912606659539.6610563982243023.96974318659727.474588227
#Sta/Elev= 30
       0 2103.93    68.7 2096.11     133 2085.44   169.7 2084.32   229.3 2085.96
   285.9 2083.72   311.9 2079.24   334.5 2070.56     354 2072.01   369.4 2069.11
   458.5 2068.67   482.9 2071.98   529.2 2074.85   599.8 2068.11   621.7 2066.45
  678.892068.109   699.5 2068.67     719 2071.32     746 2070.68   796.9 2076.65
   917.3 2075.02   999.5 2070.48  1007.7 2072.66  1018.1 2080.23  1022.3 2081.78
    1046 2080.17  1050.7 2080.93    1069 2095.93  1101.9 2106.38  1166.8 2136.64
#Mann= 6 ,-1,0
       0      .1       0   599.8    .045       0  678.89      .1       0
  731.02     .05       0  839.88     .06       0 1099.88      .1       0
#XS Ineff= 2 , 0
           526.4 2086.93  800.45         2085.03
Permanent Ineff=
       F       F
Bank Sta=599.8,678.89
XS Rating Curve= 0 ,0
Exp/Cntr(USF)=0,0
Exp/Cntr=0.3,0.1

Type RM Length L Ch R = 1 ,87339   ,337.5,337.5,337.5
XS GIS Cut Line= 3
 2242000.2330903 659388.703348972242478.09123722 659764.57089841
2242901.68649969659852.277128799
#Sta/Elev= 30
       0 2115.67    66.1 2110.88   181.9 2099.27   194.9 2097.01   240.2 2085.29
   264.6 2075.28   274.7 2068.14  279.462066.259     290 2064.01   300.2 2063.47
   371.4 2063.89  389.572066.258   396.2 2068.57   450.4 2069.87   493.6 2068.17
   529.2  2072.1   570.1 2072.97     611 2075.91     700 2073.75   753.1 2074.17
   826.2 2071.23   891.9 2071.21   912.4 2072.29   924.6 2069.58   945.1    2070
   957.3 2076.01   985.9 2076.59     990 2078.56  1002.2 2088.98  1040.5  2102.2
#Mann= 5 ,-1,0
       0      .1       0  279.46    .045       0  389.57      .1       0
     600     .06       0 1007.97      .1       0
#XS Ineff= 2 , 0
                          613.91         2079.07
Permanent Ineff=
       F       F
Bank Sta=279.46,389.57
XS Rating Curve= 0 ,0
Exp/Cntr(USF)=0,0
Exp/Cntr=0.3,0.1

Type RM Length L Ch R = 1 ,87002   ,435.7,435.7,435.7
XS GIS Cut Line= 2
2241969.58571947659824.5289210612242851.65023893660152.514102134
#Sta/Elev= 30
       0 2098.75    55.4 2092.64    61.6 2088.02    75.3 2072.25    83.8 2064.67
    88.1 2062.93   100.9 2062.49   147.9 2062.67  155.742064.659     174 2064.88
   194.8 2067.17   226.5 2067.29   250.3 2069.97   305.8 2072.49     410 2072.03
   442.3 2074.64   481.6 2072.49   497.8 2073.72     549 2072.09   630.1 2072.63
   681.3 2070.27     724    2070   741.1 2066.84   779.5 2066.94   792.3  2073.1
   822.1 2073.81   830.7 2076.74   864.8 2084.34   892.2 2095.99   941.1 2112.56
#Mann= 7 ,-1,0
       0      .1       0    83.8    .045       0  155.74      .1       0
     430     .06       0     640     .05       0     750     .06       0
     850      .1       0
#XS Ineff= 2 , 0
                           439.8         2077.49
Permanent Ineff=
       F       F
Bank Sta=83.8,155.74
XS Rating Curve= 0 ,0
Exp/Cntr(USF)=0,0
Exp/Cntr=0.3,0.1

Type RM Length L Ch R = 1 ,86566   ,505.2,505.2,505.2
XS GIS Cut Line= 3
2241917.95474636660319.5224880522242331.32803523 660252.51089464
2242776.96748926 660360.14282364
#Sta/Elev= 30
       0 2132.94    54.9 2111.42    71.1 2098.02    75.2 2096.44    95.5 2096.69
    99.5 2094.59   111.7 2081.16   127.9 2067.51  149.522062.794   160.3 2061.04
   196.8 2061.03   237.3 2061.21  241.982062.791   253.5 2069.46   257.5 2069.84
   338.7 2069.19   407.5 2071.54   448.4 2070.77   460.8 2068.66   522.8 2069.91
     576 2067.24   666.5    2068   703.6 2066.32   724.2 2072.22     753 2072.34
   769.4 2080.01   791.2 2085.96   822.9 2097.34   872.3    2103   877.2  2105.1
#Mann= 7 ,-1,0
       0      .1       0  149.52    .045       0  241.98      .1       0
     360     .06       0  568.77     .05       0  668.77     .06       0
  768.77      .1       0
#XS Ineff= 2 , 0
                          434.71         2076.38
Permanent Ineff=
       F       F
Bank Sta=149.52,241.98
XS Rating Curve= 0 ,0
Exp/Cntr(USF)=0,0
Exp/Cntr=0.3,0.1

Type RM Length L Ch R = 1 ,86061   ,188.8,188.8,188.8
XS GIS Cut Line= 3
2241966.60295854660769.9705739042242356.10623816660770.947140634
2242578.03312621660824.484368525
#Sta/Elev= 30
       0 2105.46    41.6  2087.3    57.6 2078.39    77.6 2070.18   101.6 2070.56
   113.6 2065.86   165.6 2062.34   217.6 2062.34   228.2 2060.37   237.6 2058.41
   265.6 2057.99   301.6 2058.26   313.6 2059.87  336.892060.354   349.6 2064.44
   369.6 2066.97   381.6 2065.05   401.4 2064.87   410.1 2061.46   414.3  2061.5
   422.5 2063.33     439 2070.84   451.3 2070.21     471 2073.65   504.8 2073.57
   517.1 2079.94   527.3  2079.5   554.2  2081.7   603.5 2088.87   617.8 2089.78
#Mann= 5 ,-1,0
       0      .1       0     210     .08       0   228.2    .045       0
  336.89     .06       0   609.5      .1       0
Bank Sta=228.2,336.89
XS Rating Curve= 0 ,0
Exp/Cntr(USF)=0,0
Exp/Cntr=0.3,0.1

Type RM Length L Ch R = 1 ,85872   ,61.8,61.8,61.8
XS GIS Cut Line= 2
2241939.52074227660831.458746807 2242510.2444641661016.592302215
#Sta/Elev= 30
       0 2099.84    17.8 2092.63    34.3 2083.13    46.9 2077.65    84.4  2068.5
   148.2 2068.36   173.1  2067.2   189.9 2065.13   206.7 2065.26   244.6 2062.05
   297.2 2062.23   307.7 2061.54   315.8 2059.33   337.1 2057.46   366.5 2057.31
   383.4 2057.45  390.692059.309     402 2066.25   408.6 2068.69   420.4 2068.83
     438 2070.66   454.8 2074.72   471.7 2075.06   480.1 2073.03   488.5 2075.48
   501.1 2077.01   547.4 2079.87   557.5  2082.5   567.1 2082.67     600 2087.85
#Mann= 5 ,-1,0
       0      .1       0     250     .08       0   315.8    .045       0
  390.69     .06       0     460      .1       0
Bank Sta=315.8,390.69
XS Rating Curve= 0 ,0
Exp/Cntr(USF)=0,0
Exp/Cntr=0.3,0.1

Type RM Length L Ch R = 1 ,85810   ,169.1,169.1,169.1
XS GIS Cut Line= 2
2241937.32328453660895.6661425012242508.04700636661080.799697909
#Sta/Elev= 30
       0 2092.93     7.2 2091.31      13 2088.99    36.6 2074.65    57.4 2068.89
    78.7 2069.31   108.6  2068.6   117.8 2067.37   133.4 2063.77   170.1 2062.17
   219.4 2061.31   246.9 2061.85   255.3 2061.14   263.7 2061.78     289 2061.09
  299.982060.048   314.2 2057.67   322.6 2057.31   368.6 2057.75  373.792060.053
   384.5 2069.55   389.9 2071.34   394.1  2071.7   402.5 2070.82   431.9 2074.77
   448.7 2075.19   457.2 2074.35     474 2077.62   532.9 2079.92     600  2087.3
#Mann= 6 ,-1,0
       0      .1       0     150     .08       0     250      .1       0
  299.98    .045       0  373.79     .06       0     460      .1       0
Bank Sta=299.98,373.79
XS Rating Curve= 0 ,0
Exp/Cntr(USF)=0,0
Exp/Cntr=0.3,0.1

Type RM Length L Ch R = 1 ,85641   ,313.9,313.9,313.9
XS GIS Cut Line= 2
2241822.42186729660957.7366704412242590.54615823661365.624011039
#Sta/Elev= 30
       0 2146.79    33.7  2120.7    56.3 2105.33    65.4 2096.68    83.7 2084.96
   101.6 2076.34   122.2 2070.17   151.7 2070.33   225.7 2067.45   237.5 2063.13
   251.1 2062.14   305.9 2060.37   359.8  2061.1  372.582058.909   397.3 2056.62
   445.8 2056.94   454.52058.911   463.9 2065.21   474.2 2069.55   495.6 2070.74
   518.3 2075.36   545.5 2075.36   581.7  2077.3   672.3 2086.31     713 2094.03
   744.7 2098.34   758.3  2102.9   784.8  2103.2   817.2 2112.51   869.7 2119.29
#Mann= 6 ,-1,0
       0      .1       0  372.58    .045       0   454.5     .06       0
     510      .1       0     590     .06       0     630      .1       0
Bank Sta=372.58,454.5
XS Rating Curve= 0 ,0
Exp/Cntr(USF)=0,0
Exp/Cntr=0.3,0.1

Type RM Length L Ch R = 1 ,85327   ,501.9,501.9,501.9
XS GIS Cut Line= 2
2241734.80755276661153.4402762962242284.36382367661637.295057026
#Sta/Elev= 30
       0 2111.13    17.8 2097.89    43.3 2084.91    54.6 2080.53    85.8 2079.28
    96.5 2073.71   108.4  2072.3     117 2067.89     134 2062.31   209.7 2061.39
   241.6 2059.69   298.4 2060.36   346.5 2057.72   374.9 2059.09  385.272056.087
   396.2 2054.08   440.1 2053.83   448.6 2054.22  453.262056.088   465.5 2067.33
   468.4 2068.87   488.3 2072.86   534.8 2078.81   544.4  2079.2   550.6 2078.02
   588.1 2080.11   609.4 2082.73   673.3 2094.23   719.9 2101.04   732.2 2101.51
#Mann= 7 ,-1,0
       0      .1       0     130     .08       0     270      .1       0
  385.27    .045       0  453.26      .1       0     460     .06       0
     570      .1       0
Bank Sta=385.27,453.26
XS Rating Curve= 0 ,0
Exp/Cntr(USF)=0,0
Exp/Cntr=0.3,0.1

Type RM Length L Ch R = 1 ,84825   ,440.6,440.6,440.6
XS GIS Cut Line= 2
2241499.86708766661353.3391600972241727.12108677661939.334709732
#Sta/Elev= 30
       0  2093.6    12.7 2085.54    38.4 2082.86    61.9 2069.61    85.6 2060.28
    95.9 2057.56   145.7 2055.22     180 2056.75   201.5 2054.28   281.4 2056.94
   284.5 2056.03  288.932052.867   291.6 2050.86   321.7 2050.62   360.2 2050.89
  368.182052.863   381.7  2054.7   432.9 2056.38   445.3  2064.6   463.2 2066.38
     476 2072.33   493.2 2078.35   510.2 2088.15   527.5 2089.19   536.1 2088.51
   553.5 2095.84   574.7 2100.27   604.8 2109.01   613.3 2112.77   628.5 2123.59
#Mann= 7 ,-1,0
       0     .08       0     190      .1       0  288.93    .045       0
  368.18      .1       0     400     .06       0     510      .1       0
     620     .06       0
Bank Sta=288.93,368.18
XS Rating Curve= 0 ,0
Exp/Cntr(USF)=0,0
Exp/Cntr=0.3,0.1

Type RM Length L Ch R = 1 ,84385   ,431.6,431.6,431.6
XS GIS Cut Line= 2
2241126.44108648661599.0667338652241359.73103412662151.855844044
#Sta/Elev= 30
       0  2087.4      11  2079.6    36.5 2078.87    45.7 2075.36    54.8 2069.47
    63.1 2066.68    80.4 2062.94   115.2 2059.95   134.2 2050.84   267.1 2053.02
   277.7 2052.41  286.882049.664     296 2047.54   340.9 2047.42  353.472049.663
   358.3 2051.49     367 2058.51     380 2059.38   384.4 2061.17   397.4 2072.32
   415.1 2078.62   430.4 2087.38   462.5 2088.29   475.5 2098.47   508.6 2110.27
   523.3 2117.16   552.5 2127.17   579.7 2127.39   592.2 2136.63     600 2139.49
#Mann= 6 ,-1,0
       0      .1       0     140     .08       0     250      .1       0
  286.88    .045       0  353.47      .1       0     360     .06       0
Bank Sta=286.88,353.47
XS Rating Curve= 0 ,0
Exp/Cntr(USF)=0,0
Exp/Cntr=0.3,0.1

Type RM Length L Ch R = 1 ,83953   ,439.8,439.8,439.8
XS GIS Cut Line= 3
2240732.28562249661773.0858000692240889.90371642662131.599545099
2241022.88885325662298.014140198
#Sta/Elev= 30
       0 2088.65     9.1 2088.22    26.3 2079.31    49.4 2071.61    83.1 2064.14
    96.2  2063.3   109.3 2060.53   158.7 2057.49     170 2055.32  188.882047.025
   198.5 2044.97   236.1 2044.67   275.4 2045.46   279.8 2045.98  281.852047.025
   288.3 2048.96   297.9 2049.41   319.1 2052.64   333.9 2056.56   376.3 2058.35
   444.9 2067.37     457 2070.59   462.7  2073.9   470.5 2079.77   472.2 2080.28
   485.4 2080.31   508.2 2078.51   590.7 2106.18   593.3 2106.74   604.7 2106.29
#Mann= 7 ,-1,0
       0      .1       0     170     .08       0  188.88    .045       0
  281.85      .1       0  401.63     .06       0  501.63     .07       0
  561.63     .06       0
Bank Sta=188.88,281.85
XS Rating Curve= 0 ,0
Exp/Cntr(USF)=0,0
Exp/Cntr=0.3,0.1

Type RM Length L Ch R = 1 ,83513   ,389,389,389
XS GIS Cut Line= 3
2240312.48874047662197.9468257052240406.47741649662197.657797262
 2240836.2830352662497.671224523
#Sta/Elev= 30
       0 2103.28    27.7 2100.14    63.7 2093.17      94 2083.52   112.1 2078.74
   135.1    2068   149.1 2057.11   161.32045.291   169.2 2042.63     198 2042.41
   222.9 2042.74  230.532045.289   237.5 2046.98     257 2047.06   267.2 2051.33
   278.7 2053.46   396.5  2056.4     418 2060.23   435.6 2065.18   442.6 2069.13
     457 2079.84   461.9 2080.99   505.7  2080.6   511.4 2082.96   515.6 2083.37
     540 2082.79   557.4 2080.95   559.5 2081.86   574.6 2094.71   618.1 2107.42
#Mann= 5 ,-1,0
       0      .1       0   161.3    .045       0  230.53      .1       0
  473.99     .08       0  573.99      .1       0
Bank Sta=161.3,230.53
XS Rating Curve= 0 ,0
Exp/Cntr(USF)=0,0
Exp/Cntr=0.3,0.1

Type RM Length L Ch R = 1 ,83124   ,346.4,346.4,346.4
XS GIS Cut Line= 3
2240166.73709848662525.7052294542240398.97079693662648.054971103
2240732.40143632662687.828671855
#Sta/Elev= 30
       0 2097.43    10.7 2092.05    19.7 2090.53    51.4 2076.07    60.4 2070.64
    78.5 2065.51    87.5 2059.03   101.1 2046.59  107.222043.467     119 2041.12
   161.9 2041.24  182.932043.467     196 2046.28   223.2 2046.34   245.8 2053.52
   340.2 2050.44   412.8 2051.88     449 2061.15   466.1 2067.15   501.4 2067.07
   513.5 2069.65   517.5 2070.82   533.6  2082.8   537.6 2084.46   549.7 2085.53
   573.9 2083.31   577.9  2086.7     586 2096.63     590 2099.73   598.3 2103.11
#Mann= 6 ,-1,0
       0      .1       0  107.22    .045       0  182.93      .1       0
  372.49     .06       0  472.49     .07       0  572.49      .1       0
Bank Sta=107.22,182.93
XS Rating Curve= 0 ,0
Exp/Cntr(USF)=0,0
Exp/Cntr=0.3,0.1

Type RM Length L Ch R = 1 ,82778   ,290.6,290.6,290.6
XS GIS Cut Line= 2
2240052.76106369662921.0206193872240730.81294675662915.007953607
#Sta/Elev= 30
       0 2122.51    15.4 2111.18    39.4  2096.3    55.4 2082.07    67.4  2073.8
    95.4 2048.16   103.4 2043.56  109.412041.977   119.4 2039.65   155.4 2039.26
   183.4 2039.86  197.342041.978   219.4 2047.16   231.4 2052.11   239.4  2052.7
   331.4 2051.96   419.4 2048.53   447.6 2048.69   459.4 2050.12   503.4  2049.7
   523.4 2053.03   543.4 2059.63   555.4 2061.87   595.4 2078.82   611.4 2080.14
   623.4 2083.18   651.4 2080.59   655.4 2082.68   663.4 2091.73   678.1 2095.58
#Mann= 6 ,-1,0
       0      .1       0  109.41    .045       0  197.34      .1       0
     350     .06       0     550      .1       0     650     .06       0
Bank Sta=109.41,197.34
XS Rating Curve= 0 ,0
Exp/Cntr(USF)=0,0
Exp/Cntr=0.3,0.1
