HEC-RAS study MIDFKRIV.prj: MIDFKRIV

--- MIDFKRIV.g01 (geometry) --- (continued)

Type RM Length L Ch R = 1 ,59696   ,430.9,430.9,430.9
XS GIS Cut Line= 2
2234222.11274197677558.2301504842234741.17498457678071.332273241
#Sta/Elev= 30
       0 2009.18    36.6 1989.23    43.1 1987.25    70.4 1985.38   105.4 1972.22
   126.6 1961.42   159.1 1950.44   177.3 1935.22   186.3 1923.94  198.23 1915.18
   214.7  1911.1   258.1 1911.63  269.161915.182   278.5 1919.63   305.8 1921.41
   331.6 1919.73   396.8 1922.22   408.2 1919.73   447.2 1923.22   458.9 1921.64
   478.7 1922.46   492.9 1927.01   514.7 1925.28   531.6 1927.62   574.9  1928.6
   584.6 1930.38   595.9 1936.29   604.7  1938.2   630.1 1934.96   729.9 1972.64
#Mann= 3 ,-1,0
       0      .1       0  198.23    .045       0  269.16      .1       0
#XS Ineff= 2 , 0
                          356.36          1929.4
Permanent Ineff=
       F       F
Bank Sta=198.23,269.16
XS Rating Curve= 0 ,0
Exp/Cntr(USF)=0,0
Exp/Cntr=0.3,0.1

Type RM Length L Ch R = 1 ,59265   ,325.7,325.7,325.7
XS GIS Cut Line= 2
2233982.56466325677970.394831217 2234557.7613811678295.846916366
#Sta/Elev= 30
       0 1985.41      30 1972.24    43.2 1964.22    66.2 1963.69    79.5 1957.52
   112.2 1952.94   139.7 1936.84   167.6 1933.19   181.1 1932.83   204.1 1929.01
   213.3 1925.35     227 1923.53   240.8 1915.63   268.4 1912.03   282.2 1909.34
   346.2 1912.03   358.4 1912.97   390.7 1921.39     420 1923.97   452.3 1925.37
     466 1923.05   493.4 1922.51   508.1 1919.91   521.2  1920.4   549.2 1928.23
   603.9 1954.68   613.7 1962.13   625.5 1963.61   645.3 1974.68   660.9 1978.12
#Mann= 4 ,-1,0
       0     .08       0      30      .1       0   268.4    .045       0
   346.2      .1       0
Bank Sta=268.4,346.2
XS Rating Curve= 0 ,0
Exp/Cntr(USF)=0,0
Exp/Cntr=0.3,0.1

Type RM Length L Ch R = 1 ,58940   ,559.7,559.7,559.7
XS GIS Cut Line= 2
2233805.64431456678178.5609522172234337.81024197 678585.57271498
#Sta/Elev= 30
       0 1970.77    26.5 1960.78    43.6 1957.86      55 1954.46      75    1954
    88.8 1946.53     114  1944.9   142.6 1935.94   243.4 1923.96   295.3 1920.64
   307.2 1917.28  316.761911.458   326.9 1909.66   346.1 1909.05   421.2 1908.58
   431.2 1909.18  440.311911.458   486.6 1913.31   497.3 1917.34   514.4 1918.88
   517.3 1919.94   526.9 1928.69   557.1 1941.69   570.6 1949.06   583.7 1951.15
   592.4 1956.87   637.7 1975.97   651.4 1984.55   662.9  1985.7     670 1988.53
#Mann= 3 ,-1,0
       0      .1       0  316.76    .045       0  440.31      .1       0
Bank Sta=316.76,440.31
XS Rating Curve= 0 ,0
Exp/Cntr(USF)=0,0
Exp/Cntr=0.3,0.1

Type RM Length L Ch R = 1 ,58380   ,499.2,499.2,499.2
XS GIS Cut Line= 2
2233399.71722567678432.9231833962233916.06220568678999.510845228
#Sta/Elev= 30
       0 1974.68    30.4 1973.46    42.2 1968.17    76.1 1959.82   108.6 1955.35
   124.8 1951.34   133.6 1952.54   153.4 1952.07   181.7 1944.41     210 1940.37
   227.6 1940.36   249.7 1938.23   323.3 1923.53   352.1 1921.53   400.8  1915.8
   446.1 1913.76   460.4 1912.23   472.11907.972     479  1906.4   509.1 1906.01
   588.6 1906.43  600.151907.973   612.3 1910.67   626.3 1916.99     648 1917.31
   665.8 1928.08   688.6 1934.59   699.9  1935.9   730.9 1951.21   766.6 1965.95
#Mann= 3 ,-1,0
       0      .1       0   472.1    .045       0  600.15      .1       0
Bank Sta=472.1,600.15
XS Rating Curve= 0 ,0
Exp/Cntr(USF)=0,0
Exp/Cntr=0.3,0.1

Type RM Length L Ch R = 1 ,57881   ,481.4,481.4,481.4
XS GIS Cut Line= 2
2233052.13996906678895.7184228492233737.68703228679317.407488316
#Sta/Elev= 30
       0 2008.72    28.2 1998.09      47  1992.6    56.3 1991.42    65.8  1987.3
      94 1979.83   109.7 1973.48   147.8 1962.85   220.8  1962.4     257  1937.7
   295.9 1908.63  301.271905.864   312.2 1901.86   347.6 1901.59   364.5 1902.28
  374.231905.863   385.1 1908.76   399.8 1907.58   436.8 1910.41   463.4 1910.36
   493.1 1908.47   556.4 1915.62   587.1 1914.19   624.6    1917     634    1916
   651.7 1918.15   690.4 1929.42   723.2 1941.27   765.8 1954.12   804.9 1970.19
#Mann= 3 ,-1,0
       0      .1       0  301.27    .045       0  374.23      .1       0
Bank Sta=301.27,374.23
XS Rating Curve= 0 ,0
Exp/Cntr(USF)=0,0
Exp/Cntr=0.3,0.1

Type RM Length L Ch R = 1 ,57399   ,492.4,492.4,492.4
XS GIS Cut Line= 4
2232985.96674987679486.9888734682233052.82292052679489.989179313
2233358.29591494679565.9159929532233705.96910332679536.777763157
#Sta/Elev= 30
       0 1986.28    14.2 1982.19    30.2 1973.56    50.3 1973.22    62.3 1970.29
    78.6  1969.5    86.9 1967.64     124 1940.64   136.3 1930.11   156.9 1908.44
  163.841903.201   173.4 1901.04   247.6  1901.5  253.911903.203   268.2 1907.31
   283.6 1909.73   375.4 1914.39   399.6  1913.2   423.7 1913.76   451.8 1910.48
   463.9 1911.25     496 1910.41     516 1912.07   556.2 1919.06   591.5 1929.45
   612.4 1934.28   656.5 1940.75   676.6 1948.47   695.2 1953.38   730.6 1959.49
#Mann= 3 ,-1,0
       0      .1       0  163.84    .045       0  253.91      .1       0
Bank Sta=163.84,253.91
XS Rating Curve= 0 ,0
Exp/Cntr(USF)=0,0
Exp/Cntr=0.3,0.1

Type RM Length L Ch R = 1 ,56907   ,386.1,386.1,386.1
XS GIS Cut Line= 3
2233107.89570247680058.4125357712233305.32371937680017.945395091
2233716.83475052679651.798740701
#Sta/Elev= 30
       0 1963.49     8.5 1962.69      37 1953.27    45.3  1949.4    58.9 1948.26
      86 1939.03   114.6 1932.31     135 1930.23   171.8 1922.46   221.1 1917.15
   232.1 1913.95   242.8 1904.18  251.981898.763   257.9 1897.03   296.4 1896.06
   331.6 1896.91   342.9 1898.61   362.8 1896.46  380.471898.765   401.3 1905.67
   443.4 1905.34   461.4  1909.1   478.9 1906.89   493.1 1906.95   510.5 1910.83
   527.6 1912.87   605.9 1919.24   649.7 1938.19   702.1 1946.93   752.4 1951.53
#Mann= 3 ,-1,0
       0      .1       0  251.98    .045       0  380.47      .1       0
Bank Sta=251.98,380.47
XS Rating Curve= 0 ,0
Exp/Cntr(USF)=0,0
Exp/Cntr=0.3,0.1

Type RM Length L Ch R = 1 ,56521   ,373.5,373.5,373.5
XS GIS Cut Line= 2
2233271.02087511680292.3448974772233977.30089889680186.856725623
#Sta/Elev= 30
       0 1936.82    84.7 1917.24    94.2 1916.57   126.5 1910.65   183.2 1909.41
   199.3 1906.84   211.5 1902.12   235.7 1900.48   284.3 1900.75  301.551896.662
   320.7 1894.31   348.6  1893.7   413.7 1894.92  428.961896.662     446 1904.78
   462.2 1905.18   478.4 1907.12   490.5 1916.25   494.6 1916.82   502.7 1914.76
   506.7 1915.17   518.8 1921.66     535 1925.21   547.2 1930.33   567.4  1935.9
   591.6 1938.88   611.9 1947.17   644.2 1957.19   661.8 1963.75   714.1    1979
#Mann= 3 ,-1,0
       0      .1       0  301.55    .045       0  428.96      .1       0
Bank Sta=301.55,428.96
XS Rating Curve= 0 ,0
Exp/Cntr(USF)=0,0
Exp/Cntr=0.3,0.1

Type RM Length L Ch R = 1 ,56147   ,417.5,417.5,417.5
XS GIS Cut Line= 2
2233274.54012965680456.0110775092233826.31398773680691.692238264
#Sta/Elev= 30
       0 1933.93     6.1 1933.07    14.3 1929.53    29.6 1925.01    45.3    1918
    72.2 1909.06    84.4    1906   110.5    1905   145.4 1907.46   203.3 1905.26
     228 1903.69   249.7 1900.88   267.1 1900.32   280.2 1898.11   293.2 1898.55
  300.631894.669   306.3 1892.09     313 1891.96   375.8 1892.09   384.5 1892.47
  390.241894.674   401.9 1905.65   404.4 1907.17   423.7 1909.19   431.9 1912.37
   445.4 1920.65   467.2 1926.85   493.3 1930.71   550.7 1943.49     600 1958.81
#Mann= 3 ,-1,0
       0      .1       0  300.63    .045       0  390.24      .1       0
Bank Sta=300.63,390.24
XS Rating Curve= 0 ,0
Exp/Cntr(USF)=0,0
Exp/Cntr=0.3,0.1

Type RM Length L Ch R = 1 ,55730   ,506.4,506.4,506.4
XS GIS Cut Line= 2
2233094.23463012680716.3588453042233579.53049606681069.187305748
#Sta/Elev= 30
       0 1956.56    22.2 1947.04    46.9 1938.18    53.5 1934.17    56.8 1933.14
    67.8 1932.03    76.4 1927.15    86.5 1924.17    99.3 1917.99   135.9 1903.82
   156.6 1900.05   170.9 1901.84  192.641892.948   200.2 1890.38   212.3    1890
   296.9 1890.71  305.741892.945   338.7 1898.25   357.1  1905.7   363.4 1906.93
   383.2 1904.63   395.9 1904.06   414.3 1905.33   457.4 1910.43   487.1 1917.04
   496.9 1920.35   511.8 1921.89   546.4 1929.49   583.3 1938.88     600 1944.01
#Mann= 3 ,-1,0
       0      .1       0  192.64    .045       0  305.74      .1       0
Bank Sta=192.64,305.74
XS Rating Curve= 0 ,0
Exp/Cntr(USF)=0,0
Exp/Cntr=0.3,0.1

Type RM Length L Ch R = 1 ,55223   ,532.2,532.2,532.2
XS GIS Cut Line= 2
2232787.27959156681084.9952346782233251.26101406681465.417683511
#Sta/Elev= 30
       0 1943.88    12.9 1938.73      27 1931.23    54.8 1920.12    63.2 1915.54
    77.5 1912.87    88.9  1908.6   111.6 1903.47   120.1 1902.03     140 1901.59
   213.2 1901.45   228.8 1899.75   242.4 1894.03   256.6 1893.96  267.151890.559
   279.3  1887.8   315.7 1887.51   347.5  1887.9   358.1 1890.58   373.6  1897.3
   395.8 1898.12   404.6 1901.46   429.3  1903.8   466.9 1912.16   478.3 1915.48
   506.7 1920.33   517.6 1924.52   544.3 1930.91     565 1937.34     600 1946.12
#Mann= 3 ,-1,0
       0      .1       0  267.15    .045       0   358.1      .1       0
Bank Sta=267.15,358.1
XS Rating Curve= 0 ,0
Exp/Cntr(USF)=0,0
Exp/Cntr=0.3,0.1

Type RM Length L Ch R = 1 ,54691   ,553.7,553.7,553.7
XS GIS Cut Line= 2
2232410.46826022 681451.547019172232865.37343643681842.777489164
#Sta/Elev= 30
       0 1952.84    84.6 1918.38    90.3 1915.17   100.7 1906.84   107.8 1904.17
   144.2 1902.47   158.4 1899.06   186.7  1899.5   223.3 1896.89   239.7 1897.23
   266.2 1894.44  282.681891.354   324.1 1888.15   376.8 1887.87   392.7 1887.88
  399.411891.358   422.2 1897.87   450.5 1900.07   456.2 1903.24   464.7 1906.03
   476.1 1907.66   487.1 1911.68     514 1918.63   519.3 1920.69   524.6 1924.42
   529.8 1926.25     547 1925.07   561.5 1926.48     581 1935.06     600 1941.18
#Mann= 3 ,-1,0
       0      .1       0  282.68    .045       0  399.41      .1       0
Bank Sta=282.68,399.41
XS Rating Curve= 0 ,0
Exp/Cntr(USF)=0,0
Exp/Cntr=0.3,0.1

Type RM Length L Ch R = 1 ,54138   ,731.2,731.2,731.2
XS GIS Cut Line= 2
2232016.43785499681769.4114677372232501.05412835682255.028714403
#Sta/Elev= 30
       0  1945.2    16.6 1939.47    67.5 1926.08   126.9  1907.6   143.9 1905.78
   163.8 1902.04   203.1 1899.13   214.6 1897.31   240.1 1895.37   254.2 1891.93
   259.9 1891.73   268.4 1893.58   282.2 1894.32   296.6 1892.93  305.721889.551
   310.5 1887.83   316.4 1887.28   389.6 1887.12   421.1 1887.55  432.94 1889.55
   446.1 1893.26   500.3 1896.19   573.8 1903.96   585.1 1906.86   594.2 1910.66
   616.2 1910.16   628.2 1915.25   650.8  1919.4   675.6 1922.45   686.1 1925.61
#Mann= 3 ,-1,0
       0      .1       0  305.72    .045       0  432.94      .1       0
#XS Ineff= 2 , 0
          279.76 1901.72
Permanent Ineff=
       F       F
Bank Sta=305.72,432.94
XS Rating Curve= 0 ,0
Exp/Cntr(USF)=0,0
Exp/Cntr=0.3,0.1

Type RM Length L Ch R = 1 ,53406   ,751.7,751.7,751.7
XS GIS Cut Line= 2
2231555.79978446682121.6795394022231948.81436603682809.813245151
#Sta/Elev= 30
       0 1962.01    43.9 1932.18    57.2  1929.9    81.4 1916.54   155.3 1887.42
   179.1 1884.75   183.7 1885.43   193.4 1891.26   202.2 1893.59   249.1 1893.41
   266.7 1895.41   294.2 1895.51   418.6 1892.19   436.3 1889.05   473.21886.648
   510.1 1883.47   565.3 1883.73   570.6 1886.62   579.8 1898.91   584.4 1901.23
     589  1902.2   612.7 1899.12   621.5 1900.03   630.3 1904.53   639.7 1912.66
   644.3 1914.94   706.5 1935.06   762.2 1958.09   782.5 1960.58   792.5 1966.73
#Mann= 3 ,-1,0
       0      .1       0   473.2    .045       0   570.6      .1       0
Bank Sta=473.2,570.6
XS Rating Curve= 0 ,0
Exp/Cntr(USF)=0,0
Exp/Cntr=0.3,0.1

Type RM Length L Ch R = 1 ,52655   ,626.1,626.1,626.1
XS GIS Cut Line= 2
2231113.28921326682264.0475345882231117.73834006683004.146069181
#Sta/Elev= 30
       0 1961.56     5.1 1960.86    37.1 1947.03    49.1 1938.17    61.1 1936.23
    77.1 1923.81   137.1 1892.33   169.1 1883.11   181.1 1883.36   193.1 1887.59
   202.8 1889.04   289.1 1888.31   385.1 1894.25   397.1 1892.69   417.1 1893.95
   445.1 1892.97   493.1 1887.15  511.111883.632   521.4 1881.19   552.7 1880.89
   601.1 1881.23  605.681883.681   613.1 1891.58   617.1 1894.01   633.1 1895.32
   649.1 1905.01   685.1 1914.45   705.1 1918.14   713.1 1921.96   740.1 1930.46
#Mann= 4 ,-1,0
       0      .1       0  511.11    .045       0  605.68      .1       0
     730     .08       0
Bank Sta=511.11,605.68
XS Rating Curve= 0 ,0
Exp/Cntr(USF)=0,0
Exp/Cntr=0.3,0.1

Type RM Length L Ch R = 1 ,52028   ,492.2,492.2,492.2
XS GIS Cut Line= 2
 2230634.2356678682222.3453995362230473.61857503682894.057625379
#Sta/Elev= 30
       0 1937.82       7 1936.08    15.3 1931.58    31.7 1929.98    77.1 1914.36
   105.7 1900.53   118.1 1899.56   142.7 1893.42   175.6 1892.39     188 1893.45
     225 1882.67     243    1884   257.9 1881.61   270.2 1883.41  283.661881.088
     299 1878.69   356.6 1878.43     399 1878.62  409.441881.086   430.6 1886.48
   447.1 1886.69   459.4 1889.95   508.8    1891   521.1 1894.99     554 1896.84
   611.6 1903.55   632.2 1903.33   640.4 1906.76     661 1911.06   690.6 1919.94
#Mann= 5 ,-1,0
       0      .1       0  283.66    .045       0  409.44      .1       0
     590     .08       0     690      .1       0
Bank Sta=283.66,409.44
XS Rating Curve= 0 ,0
Exp/Cntr(USF)=0,0
Exp/Cntr=0.3,0.1

Type RM Length L Ch R = 1 ,51536   ,513.6,513.6,513.6
XS GIS Cut Line= 2
2230249.41877858681989.4863686512229959.04727191682731.726624696
#Sta/Elev= 30
       0 1946.61    93.3 1927.88   137.1 1920.14     152 1918.92   240.2  1901.6
   253.1 1896.79   278.9 1899.13   287.8 1896.12   315.6 1891.54   330.4  1882.4
   340.3 1879.14   351.9 1876.92   433.5 1876.83   446.4 1877.29  453.151879.194
   476.4 1882.03   562.3 1881.32     575 1880.51   588.1 1876.46   618.2 1875.91
   631.1 1877.61   639.7 1881.55   648.2  1888.4   652.5 1890.14   678.3 1889.89
   689.2 1894.23     717 1896.59   751.3 1897.31   785.7 1910.91     797 1919.62
#Mann= 4 ,-1,0
       0      .1       0   340.3    .045       0  453.15      .1       0
     760     .08       0
Bank Sta=340.3,453.15
XS Rating Curve= 0 ,0
Exp/Cntr(USF)=0,0
Exp/Cntr=0.3,0.1

Type RM Length L Ch R = 1 ,51023   ,555.3,555.3,555.3
XS GIS Cut Line= 3
2229842.00600493681765.0889116682229745.59217754681893.161118022
2229508.68034005682519.103179565
#Sta/Elev= 30
       0 1956.86    70.2 1923.87    95.2  1914.4   105.3 1908.52   140.3 1905.38
   168.9 1894.58   251.4 1892.31   292.9 1888.46   331.4 1887.39   348.5 1882.97
   366.2 1881.89   378.1 1876.53   382.7 1874.64   391.3 1874.09   528.1 1874.06
  541.63 1876.56   549.5 1880.29   567.9 1880.74   596.6 1877.66     618 1878.55
   652.2 1873.53   677.8  1874.2   690.7 1878.37     712 1878.36   724.9 1884.76
     742 1886.09   759.1 1899.34   784.8  1911.5   811.6 1926.64   829.6 1934.12
#Mann= 3 ,-1,0
       0      .1       0   378.1    .045       0  541.63      .1       0
Bank Sta=378.1,541.63
XS Rating Curve= 0 ,0
Exp/Cntr(USF)=0,0
Exp/Cntr=0.3,0.1

Type RM Length L Ch R = 1 ,50467   ,47.3,47.3,47.3
XS GIS Cut Line= 4
2228933.95703236 682059.025500692229076.56215578682160.723964817
2229205.71619273 682486.000080182229398.32546388682647.792709999
#Sta/Elev= 30
       0 1925.96      42 1913.78    86.2 1905.47     103 1900.12   127.7 1899.99
   160.9 1889.17   175.2 1887.62   184.3 1888.23   199.9 1876.59   210.1 1872.64
   282.5 1872.09   295.3 1876.59     322 1882.83   347.5 1883.03     360 1876.55
   369.3 1875.84   378.5 1877.19   395.1 1882.89   433.9 1885.09   442.5 1889.06
   459.7 1889.29   472.6 1885.34   498.4 1885.74   507.9 1887.78     521 1894.74
   536.3 1896.43   622.4 1898.69   685.5 1903.83   747.7 1905.19   776.7 1908.23
#Mann= 5 ,-1,0
       0      .1       0      70     .06       0  195.15      .1       0
   199.9    .045       0   295.3     .06       0
Bank Sta=199.9,295.3
XS Rating Curve= 0 ,0
Exp/Cntr(USF)=0,0
Exp/Cntr=0.3,0.1

Type RM Length L Ch R = 1 ,50420   ,524.1,524.1,524.1
XS GIS Cut Line= 4
2228889.20571361682073.0400840162229031.81083703682174.738548144
2229173.60773533682520.5593131932229374.11879481682668.128723998
#Sta/Elev= 30
       0 1937.81     5.1 1936.66    16.6 1930.04    42.4 1919.37    65.3 1911.41
   103.6 1906.75   116.9 1902.53     138 1902.91   155.9 1899.19   171.4 1892.18
   186.3 1887.83   195.7 1881.66   215.6 1876.31   229.4 1872.71   239.4 1872.32
   285.9 1873.46  295.07 1876.37   302.6 1878.33   330.6 1880.95   398.8 1881.29
     528 1886.01     550 1892.91   556.9 1893.23   562.6 1891.89     572 1894.62
   588.4 1894.93   601.8 1897.29     716 1901.36     760 1906.21   797.9 1908.14
#Mann= 6 ,-1,0
       0      .1       0     120     .06       0   215.6    .045       0
  295.07     .06       0  668.92      .1       0  688.92     .06       0
Bank Sta=215.6,295.07
XS Rating Curve= 0 ,0
Exp/Cntr(USF)=0,0
Exp/Cntr=0.3,0.1

Type RM Length L Ch R = 1 ,49896   ,413.3,413.3,413.3
XS GIS Cut Line= 2
2228599.16010338 682679.262134632229489.60603593 682716.96768049
#Sta/Elev= 30
       0 2010.23    53.1 1976.73    89.1 1951.53   101.1 1942.82   109.1 1931.18
   125.1 1926.78   145.1  1908.9     168 1891.41   185.2 1883.26   205.2 1879.91
   216.4 1875.81   229.2 1871.28  258.171875.788   291.7 1881.77   309.3 1879.99
   325.3 1875.89   344.7 1878.43     360 1877.76   393.4 1886.26   425.4 1886.88
   449.4 1880.41   477.4 1884.24   521.5 1882.78   541.5 1891.44   546.7 1892.14
   581.5 1891.61   621.6 1894.74   694.2 1896.86   853.8 1916.84   891.2 1918.19
#Mann= 6 ,-1,0
       0      .1       0   216.4    .045       0  258.17      .1       0
     290     .12       0     490      .1       0     790     .06       0
Bank Sta=216.4,258.17
XS Rating Curve= 0 ,0
Exp/Cntr(USF)=0,0
Exp/Cntr=0.3,0.1

Type RM Length L Ch R = 1 ,49483   ,385.4,385.4,385.4
XS GIS Cut Line= 3
2228813.15724026683216.1877963462229321.69031766682785.347272433
2229507.30990183682732.688903765
#Sta/Elev= 30
       0 1972.56      17 1959.75    35.4  1948.7    72.7 1935.39    95.1 1930.98
   108.8 1923.39   134.8 1920.42   165.5 1901.26   188.8 1893.52  223.771874.573
   234.2 1871.02   245.1 1870.66     308 1872.87  316.42 1874.57   326.4 1880.24
   353.4 1886.54   378.9 1885.93   394.5 1878.82   402.4 1877.16   432.8 1877.06
   439.1 1878.62   449.6 1884.43   466.9 1884.88   486.3 1889.69   557.7 1888.64
   617.7 1894.87   684.8 1897.81   810.5 1914.37   837.1  1920.5   859.4 1920.19
#Mann= 4 ,-1,0
       0      .1       0  223.77    .045       0  316.42      .1       0
  726.51     .06       0
Bank Sta=223.77,316.42
XS Rating Curve= 0 ,0
Exp/Cntr(USF)=0,0
Exp/Cntr=0.3,0.1

Type RM Length L Ch R = 1 ,49097   ,524.2,524.2,524.2
XS GIS Cut Line= 2
2229114.52079033683560.3398163232229576.66564916682924.753786791
#Sta/Elev= 30
       0 1964.93    29.2 1950.76   112.3 1922.55   137.4 1911.31   149.5 1910.08
   172.1 1901.14     182 1900.41   215.3 1893.42   232.5 1892.72   280.9 1886.51
   290.8 1883.19  307.441872.729   315.5 1870.23   329.3 1869.88   399.6 1870.01
  417.931872.727   438.1 1875.08   444.4 1878.54   463.9 1884.39   493.5 1883.99
   503.4 1884.71   513.3 1887.11   552.9 1885.49   567.6 1886.52   601.4 1885.67
     632 1884.03   686.4 1885.08   701.2 1888.33   750.8 1905.93   785.8 1913.96
#Mann= 3 ,-1,0
       0      .1       0  307.44    .045       0  417.93      .1       0
Bank Sta=307.44,417.93
XS Rating Curve= 0 ,0
Exp/Cntr(USF)=0,0
Exp/Cntr=0.3,0.1

Type RM Length L Ch R = 1 ,48573   ,605.9,605.9,605.9
XS GIS Cut Line= 2
 2229344.2935005683767.8440107042230012.87747543683337.737714092
#Sta/Elev= 30
       0 1935.56    53.9 1915.38    66.4 1910.05    77.1 1903.37    94.5 1900.06
   118.8 1890.41   142.5 1886.53   218.6 1881.19   300.7 1881.82   359.8 1875.79
   401.3 1875.44  436.31 1870.38   456.2 1867.69   499.7 1867.28   529.9 1867.51
  550.651870.378     572 1875.28   580.1 1883.06   584.9 1885.29   599.1 1883.53
   608.7 1884.48   644.4 1905.27   656.2 1910.87   670.5 1912.62   699.4 1923.44
   714.7  1929.9   728.3 1937.87   756.1 1939.74     763 1944.15     795 1957.15
#Mann= 5 ,-1,0
       0      .1       0  436.31    .045       0  550.65      .1       0
     720     .06       0     750      .1       0
Bank Sta=436.31,550.65
XS Rating Curve= 0 ,0
Exp/Cntr(USF)=0,0
Exp/Cntr=0.3,0.1

Type RM Length L Ch R = 1 ,47967   ,483.6,483.6,483.6
XS GIS Cut Line= 2
2229496.96022196684019.7304303972230096.61600319684040.051454832
#Sta/Elev= 30
       0 1909.85    51.2 1894.67    63.3 1887.47    79.3 1887.78    95.3 1883.11
   111.3 1879.94   191.3 1877.68   251.4 1879.82   287.4 1878.11   307.4 1878.49
   316.7 1876.17  333.331868.645   347.4 1865.54   379.4  1864.5   419.5 1864.79
  435.011868.643   451.5 1875.93   467.5 1889.22   475.5 1891.22   487.5 1890.41
   499.5 1891.99   515.5 1904.84   527.5 1918.18   539.5 1920.41   555.5 1932.05
   559.5 1933.56   567.5 1934.26   571.5 1936.27   575.5 1939.69     600 1950.86
#Mann= 3 ,-1,0
       0      .1       0  333.33    .045       0  435.01      .1       0
#XS Ineff= 2 , 0
          250.31 1886.51
Permanent Ineff=
       F       F
Bank Sta=333.33,435.01
XS Rating Curve= 0 ,0
Exp/Cntr(USF)=0,0
Exp/Cntr=0.3,0.1

Type RM Length L Ch R = 1 ,47484   ,495.4,495.4,495.4
XS GIS Cut Line= 2
2229431.31588691684252.4976893422229923.88509187684595.098883627
#Sta/Elev= 30
       0 1911.89    29.2 1901.47      40 1895.75    55.7 1895.15    70.1 1890.16
   116.1 1881.34   176.3 1874.69   193.6 1875.44   215.4 1873.79     231 1874.51
   259.3  1871.4  272.231866.878   283.6 1863.58   312.9 1862.95   340.2 1864.45
  359.711866.878   377.6 1869.44   389.1 1872.58   393.5 1874.93   407.5 1886.05
   414.5 1887.73   428.5 1887.96   432.2 1889.01   449.5 1901.79   460.9 1907.72
   533.6 1933.11   547.1 1939.47   561.5 1941.06     573 1946.83     600 1955.05
#Mann= 3 ,-1,0
       0      .1       0  272.23    .045       0  359.71      .1       0
Bank Sta=272.23,359.71
XS Rating Curve= 0 ,0
Exp/Cntr(USF)=0,0
Exp/Cntr=0.3,0.1

Type RM Length L Ch R = 1 ,46988   ,414.7,414.7,414.7
XS GIS Cut Line= 2
2229077.67825458684476.0613978692229510.08245632684892.026067423
#Sta/Elev= 30
       0  1973.4       9 1969.57    20.1  1966.8    64.8 1945.85    70.1  1941.6
    76.6  1934.7    90.3 1932.47   111.2 1914.87     127 1913.43   132.7 1911.57
   168.9 1890.05   192.2 1880.21   197.8 1876.19  207.981866.376   214.4 1862.81
   219.9 1861.87   301.6 1861.14   316.6 1862.97  332.091866.378     342 1868.19
   382.4 1870.86   399.7 1875.15   426.9 1875.14   460.8 1877.11   480.7 1880.94
     503 1880.29   508.9 1881.89   559.9 1888.36   586.3 1894.13     600  1898.4
#Mann= 3 ,-1,0
       0      .1       0  207.98    .045       0  332.09      .1       0
Bank Sta=207.98,332.09
XS Rating Curve= 0 ,0
Exp/Cntr(USF)=0,0
Exp/Cntr=0.3,0.1

Type RM Length L Ch R = 1 ,46573   ,510.4,510.4,510.4
XS GIS Cut Line= 2
2228839.23968153684862.2189102682229329.00784081685208.812548627
#Sta/Elev= 30
       0 1940.22    45.2 1915.04    60.2 1913.97    74.6 1905.61   117.6 1888.43
   143.3 1880.45   148.2 1877.14  158.021866.013   162.9 1862.28   167.8 1860.94
   221.7  1862.9   260.9 1860.85   268.3 1862.49  276.711866.014   286.9 1869.91
   302.9 1871.82   329.9 1869.44   334.4 1869.97   352.9 1875.43   388.3 1874.25
   406.7 1876.82   427.5 1877.53   436.1 1880.62   466.7 1888.04   505.9 1899.97
   520.6 1905.36   533.7 1908.51   579.9  1925.7   591.1 1931.15     600 1932.22
#Mann= 3 ,-1,0
       0      .1       0  158.02    .045       0  276.71      .1       0
Bank Sta=158.02,276.71
XS Rating Curve= 0 ,0
Exp/Cntr(USF)=0,0
Exp/Cntr=0.3,0.1

Type RM Length L Ch R = 1 ,46063   ,485.1,485.1,485.1
XS GIS Cut Line= 2
2228528.48195682 685269.24117084 2229034.6841574685591.358124956
#Sta/Elev= 30
       0 1908.18    14.2 1901.48    31.6 1901.09    43.2 1895.52   106.9 1880.03
   146.6 1875.91   160.8 1875.17   184.5  1875.9  216.881865.866   231.5 1860.97
     246 1858.57   288.8  1859.5   331.5 1858.88   338.2 1860.64  348.411865.871
   356.1 1871.27   364.7 1874.33   376.4 1875.45   399.6 1875.25   408.3 1877.07
   424.6 1878.07     450 1883.32   473.8 1891.52   506.9 1908.27   528.9 1917.56
   549.6 1924.21   559.1 1925.52   568.6  1930.8   587.5 1939.12     600 1943.14
#Mann= 3 ,-1,0
       0      .1       0  216.88    .045       0  348.41      .1       0
Bank Sta=216.88,348.41
XS Rating Curve= 0 ,0
Exp/Cntr(USF)=0,0
Exp/Cntr=0.3,0.1

Type RM Length L Ch R = 1 ,45578   ,565.1,565.1,565.1
XS GIS Cut Line= 3
2228291.60534669  685733.83395482228774.31096351685864.797574496
2228925.48867017685853.567382492
#Sta/Elev= 30
       0 1927.05      13  1919.9    29.6 1918.07    48.8 1909.82   100.1 1892.97
   116.6 1886.17   129.1 1883.76   141.5 1876.99   145.7 1873.87   149.8 1869.51
  156.251864.858   166.4 1858.75  208.711864.858   247.7 1870.54   282.4 1868.38
     299 1868.54     328  1874.4   340.4 1875.57     410 1875.39   427.5 1873.53
   435.8 1873.94   444.1 1876.02   473.1 1875.31   485.5    1881   493.8 1882.36
     510 1887.23   542.6 1900.02   614.3 1913.89   634.4 1916.02   651.8 1922.21
#Mann= 3 ,-1,0
       0      .1       0  156.25    .045       0  208.71      .1       0
Bank Sta=156.25,208.71
XS Rating Curve= 0 ,0
Exp/Cntr(USF)=0,0
Exp/Cntr=0.3,0.1

Type RM Length L Ch R = 1 ,45013   ,478.9,478.9,478.9
XS GIS Cut Line= 2
2228530.51271135686429.4288578132228930.77655177685942.665594429
#Sta/Elev= 30
       0 1935.56    15.9 1932.88    31.4  1925.1      44 1923.91    58.2 1917.09
    63.9 1917.09    90.8 1922.09   103.9 1922.06   114.3 1919.75   137.8 1907.78
   149.1 1900.64   160.1 1891.34   174.7 1876.37  193.47 1861.64   197.4 1859.37
   202.3 1858.43   233.4 1858.27   274.2 1859.14  281.421861.638   290.3 1866.55
   300.7 1870.16   323.8 1874.24   402.1 1873.91   436.2 1871.02   478.8 1874.59
   504.4 1874.84   512.7 1877.04   544.2 1881.57   598.1  1902.3   630.2 1909.77
#Mann= 3 ,-1,0
       0      .1       0  193.47    .045       0  281.42      .1       0
Bank Sta=193.47,281.42
XS Rating Curve= 0 ,0
Exp/Cntr(USF)=0,0
Exp/Cntr=0.3,0.1

Type RM Length L Ch R = 1 ,44534   ,436.8,436.8,436.8
XS GIS Cut Line= 3
 2229027.6246349  686635.3877168 2229099.2070963686461.617644506
2229188.63236391686025.927098761
#Sta/Elev= 30
       0 1930.38    81.8 1907.28    93.2 1902.98   110.5 1899.71   132.2 1892.14
   145.1 1891.13   158.4 1886.55   200.6 1876.91   212.9 1871.52   221.1 1865.65
  231.671859.991   237.4 1857.22   241.5 1856.86   290.8 1856.66   335.4 1857.79
  344.481859.993   351.7    1864   368.1 1868.98   384.4 1871.22   421.1  1871.4
   449.7 1869.83   457.9 1873.04   466.1 1874.06   474.2 1873.64   482.4 1870.66
   486.5    1871   498.7 1878.15   600.8 1913.68   612.6 1920.57   632.7 1922.73
#Mann= 3 ,-1,0
       0      .1       0  231.67    .045       0  344.48      .1       0
Bank Sta=231.67,344.48
XS Rating Curve= 0 ,0
Exp/Cntr(USF)=0,0
Exp/Cntr=0.3,0.1

Type RM Length L Ch R = 1 ,44097   ,402.5,402.5,402.5
XS GIS Cut Line= 2
2229363.20742236686804.8077539872229676.16855884 686144.91221422
#Sta/Elev= 30
       0  1912.1    39.6 1902.72   123.5  1885.5   145.7 1882.69   154.5 1880.24
   170.3 1880.41   234.2 1873.31   331.6 1867.41   384.8 1861.93   389.2 1861.06
  391.771859.468     398 1856.51   406.9 1854.59   495.4 1855.31   499.8    1857
  503.431859.469   508.7 1862.95   516.9 1871.32     522 1875.18   539.7 1880.81
   557.4 1897.54   586.6 1916.06   599.7 1922.97   610.5 1930.41   627.7 1939.55
   645.9 1953.17   663.6 1955.01   673.1  1963.3   703.1 1979.67   730.3    1993
#Mann= 5 ,-1,0
       0      .1       0  391.77    .045       0  503.43      .1       0
     530     .06       0     730      .1       0
Bank Sta=391.77,503.43
XS Rating Curve= 0 ,0
Exp/Cntr(USF)=0,0
Exp/Cntr=0.3,0.1

Type RM Length L Ch R = 1 ,43695   ,433.1,433.1,433.1
XS GIS Cut Line= 2
2229555.61295986686977.7961951472230088.39433939686420.449441653
#Sta/Elev= 30
       0 1913.69     114 1886.89   147.9 1883.18   193.2 1875.27   267.1 1870.41
     363 1867.64   377.1 1865.41   392.31858.732   399.7 1854.72   416.7 1857.34
   463.9 1854.44   484.6 1855.21   491.81858.732   498.8 1864.43   504.4 1871.23
   509.9 1874.79   526.5 1875.43   532.1 1877.36   559.7 1900.78   568.1 1906.24
   609.1 1924.29   628.9 1936.38   631.8 1937.45   649.2 1938.25     660 1947.78
   666.5 1951.39   682.7 1958.16   709.2 1971.27   731.3 1983.56     771 2001.18
#Mann= 5 ,-1,0
       0      .1       0   392.3    .045       0   491.8      .1       0
     630     .06       0     760      .1       0
Bank Sta=392.3,491.8
XS Rating Curve= 0 ,0
Exp/Cntr(USF)=0,0
Exp/Cntr=0.3,0.1

Type RM Length L Ch R = 1 ,43261   ,414.3,414.3,414.3
XS GIS Cut Line= 2
2229753.65000275687192.5805180182230394.45617011 686761.35466318
#Sta/Elev= 30
       0 1917.57    99.5 1891.84   119.5  1884.6   133.2  1884.2   149.4 1878.83
   185.2 1872.51   257.9  1866.6   292.5 1867.66   315.5 1866.07   335.7 1867.38
   355.9 1863.52   396.2 1861.68  404.191857.055     408 1854.26   412.9 1853.84
   485.2 1854.06  492.391857.061     500 1864.16   509.3 1871.76   528.8 1873.33
     549 1889.97   580.7 1902.43   591.3 1908.11   612.4 1909.17   652.7 1926.91
   673.2  1937.5   682.9 1940.39     707 1942.85   721.4 1952.29   772.4  1974.4
#Mann= 5 ,-1,0
       0      .1       0  404.19    .045       0  492.39      .1       0
     500     .06       0     620      .1       0
Bank Sta=404.19,492.39
XS Rating Curve= 0 ,0
Exp/Cntr(USF)=0,0
Exp/Cntr=0.3,0.1

Type RM Length L Ch R = 1 ,42847   ,487.7,487.7,487.7
XS GIS Cut Line= 2
2229990.78880794687459.0636609622230593.87832052687082.871795995
#Sta/Elev= 30
       0 1896.56     8.2 1891.57    31.4 1887.29    41.4 1882.81      64 1875.32
   114.8 1870.12   162.1 1869.53   179.5 1865.54  194.15 1856.81   199.8 1853.61
   211.4 1851.81     321 1852.48  336.711856.813   359.9 1860.85   388.2 1863.19
   407.1  1868.1   423.4 1868.38   506.1 1874.12   525.1 1876.17   547.7 1880.59
   559.8 1881.73   567.4 1880.98   581.5 1888.73   593.1 1890.82   609.8 1896.92
   623.3 1900.12     644 1909.04   664.3 1913.21   693.4 1925.32   710.8 1930.32
#Mann= 5 ,-1,0
       0      .1       0  194.15    .045       0  336.71      .1       0
     460     .06       0     680      .1       0
Bank Sta=194.15,336.71
XS Rating Curve= 0 ,0
Exp/Cntr(USF)=0,0
Exp/Cntr=0.3,0.1

Type RM Length L Ch R = 1 ,42359   ,477.7,477.7,477.7
XS GIS Cut Line= 2
2230247.64253696687838.2841952432230891.13759356 687453.82714321
#Sta/Elev= 30
       0 1919.25    50.8 1897.74    65.4 1894.97    79.8 1889.29   123.7 1876.94
   135.7 1871.84   154.4  1867.6     185  1868.1   196.6  1864.9   208.3 1858.82
  219.341856.458   238.3 1851.73   330.8  1852.8   336.1 1854.13  338.851856.461
   345.4  1861.1   368.7 1861.22   377.5  1868.2   382.7 1869.19     420 1869.97
     434 1865.46   452.6 1864.68   503.8  1866.9   559.8 1873.61   615.7 1875.65
   634.2 1882.48   657.6 1893.79   672.1 1894.58   680.9 1899.23   749.6  1921.8
#Mann= 5 ,-1,0
       0      .1       0  219.34    .045       0  338.85      .1       0
     370     .06       0     450      .1       0
#XS Ineff= 2 , 0
                          418.32         1876.83
Permanent Ineff=
       F       F
Bank Sta=219.34,338.85
XS Rating Curve= 0 ,0
Exp/Cntr(USF)=0,0
Exp/Cntr=0.3,0.1

Type RM Length L Ch R = 1 ,41882   ,560.4,560.4,560.4
XS GIS Cut Line= 2
2230552.75492329  688193.85172532231196.88337735687815.206101039
#Sta/Elev= 30
       0 1897.17      55 1880.68      79  1874.3   108.2 1868.13   119.9 1864.13
   129.2 1862.57   152.4 1862.48   157.9 1860.45  164.961855.485   169.6 1852.19
     175  1851.2   268.9 1850.63   289.4 1855.54   300.9 1857.44   333.2 1855.89
   347.3 1860.29   356.6 1861.69   407.6  1859.4   426.2 1862.22   444.8 1863.19
   449.4 1864.61     454 1868.16   458.7 1869.85   477.2 1867.79   514.4 1866.87
     570  1867.7   593.3 1869.03     700  1894.5   719.6 1900.81   747.2 1905.72
#Mann= 4 ,-1,0
       0      .1       0  164.96    .045       0   289.4     .06       0
     380      .1       0
Bank Sta=164.96,289.4
XS Rating Curve= 0 ,0
Exp/Cntr(USF)=0,0
Exp/Cntr=0.3,0.1

Type RM Length L Ch R = 1 ,41321   ,345.1,345.1,345.1
XS GIS Cut Line= 3
2230810.68815931688614.5421354672231421.15500181688297.987090689
2231545.66969906 688112.49826018
#Sta/Elev= 30
       0 1901.41    96.3 1877.43   105.3 1874.27   129.7 1869.03   153.4 1866.66
   177.2 1867.14   208.9 1858.43   240.5 1858.26   258.5 1856.65     263 1855.19
   275.1 1851.26     281 1850.75   378.9 1851.21   387.8 1855.03   407.2 1855.19
   420.7 1857.11   432.4 1860.61   443.2  1866.3   454.8 1867.65   470.9  1863.2
   483.8 1863.89   509.5 1868.02     628 1868.27     673 1871.54   686.6 1874.91
   712.7 1876.04   791.3 1885.78   822.3 1891.55   862.1    1902   911.1 1908.24
#Mann= 4 ,-1,0
       0      .1       0     263    .045       0   387.8     .06       0
     500      .1       0
Bank Sta=263,387.8
XS Rating Curve= 0 ,0
Exp/Cntr(USF)=0,0
Exp/Cntr=0.3,0.1

Type RM Length L Ch R = 1 ,40976   ,509.2,509.2,509.2
XS GIS Cut Line= 4
2230797.52354856 688810.379547372230898.69219891688853.998950784
2231479.42441693688757.0794522362231721.85487744688266.047638234
#Sta/Elev= 30
       0 1923.45    42.1 1904.76    81.3  1893.2     136 1884.04   192.8 1870.95
   225.2 1866.74   290.1 1866.71  312.971854.634   322.6  1851.6   387.4 1850.55
   414.5 1854.64     432 1851.43   455.3 1850.96   472.6 1854.54   492.9 1854.32
     505  1857.6   553.7 1858.38   565.9 1860.66   618.6 1860.02     696 1864.07
   709.7 1860.19   725.6  1859.9   743.4 1862.93   801.4 1861.46   868.3 1865.29
  1037.9 1869.52  1051.2 1870.84    1078 1879.28  1197.6 1890.57  1246.6 1897.78
#Mann= 5 ,-1,0
       0      .1       0  312.97    .045       0   414.5      .1       0
  470.17     .06       0  490.17      .1       0
Bank Sta=312.97,414.5
XS Rating Curve= 0 ,0
Exp/Cntr(USF)=0,0
Exp/Cntr=0.3,0.1

Type RM Length L Ch R = 1 ,40467   ,564.5,564.5,564.5
XS GIS Cut Line= 3
2230747.69380914688881.3341227282231243.99243665689324.862911344
2231302.86732696689518.668103685
#Sta/Elev= 30
       0 1911.34    11.8 1909.28    41.8 1901.97    59.7  1896.1   127.7 1878.33
   209.9 1861.34   221.2 1861.34   263.5 1867.37     344 1870.53   381.5 1868.04
   425.2 1867.43   450.7 1863.91   483.5 1856.49   490.3 1856.01   510.3 1856.69
  531.791854.097   566.8  1849.1   578.1 1849.83  587.111854.098   595.1 1857.55
   628.3 1859.81   642.1 1865.64   655.1 1866.31   665.6 1868.68   674.3 1868.79
     691 1871.24   716.1 1877.09     783 1890.16     829 1900.81   868.2 1912.26
#Mann= 4 ,-1,0
       0      .1       0  531.79    .045       0  587.11     .06       0
     610      .1       0
#XS Ineff= 2 , 0
             342 1876.18
Permanent Ineff=
       F       F
Bank Sta=531.79,587.11
XS Rating Curve= 0 ,0
Exp/Cntr(USF)=0,0
Exp/Cntr=0.3,0.1

Type RM Length L Ch R = 1 ,39902   ,540.9,540.9,540.9
XS GIS Cut Line= 2
2230619.79811748 688889.196860962230624.17518203689594.618024492
#Sta/Elev= 30
       0  1918.4      48 1898.66      96 1874.05   112.3 1868.52     156 1864.78
     216 1866.52     256 1859.03   274.7 1857.46     296  1857.6     344 1861.78
     384 1861.22     408 1857.53  420.811851.188     436 1848.73   490.7 1847.62
     512 1848.73  524.171851.186     544 1862.24     564 1863.08     572 1868.34
     584 1868.46     600 1873.88     648 1888.11     656 1891.85     668 1893.08
     676 1898.04     700 1905.95     700 1905.97     700 1905.99   705.4 1908.52
#Mann= 5 ,-1,0
       0      .1       0  420.81    .045       0  524.17     .06       0
     600      .1       0     700     .08       0
#XS Ineff= 2 , 0
          342.79 1867.74
Permanent Ineff=
       F       F
Bank Sta=420.81,524.17
XS Rating Curve= 0 ,0
Exp/Cntr(USF)=0,0
Exp/Cntr=0.3,0.1

Type RM Length L Ch R = 1 ,39362   ,683.4,683.4,683.4
XS GIS Cut Line= 3
2230027.56515861688856.1479249422230060.94673574  688979.5626736
 2230105.7827388689737.398832584
#Sta/Elev= 30
       0 1978.88      47 1947.42    63.2  1929.6    75.7 1921.34    88.1  1908.2
   133.5 1875.58   149.5 1862.15   169.5 1853.84   257.7 1851.51     430 1854.65
  450.241849.732   470.1 1845.98   529.7 1845.96   550.2 1846.25  564.171849.732
   586.3 1858.81   598.3 1859.84   622.3 1857.75   642.4  1866.4   658.4 1868.92
   678.4 1881.02   698.5 1887.93   718.5 1891.02   750.6 1892.63   762.6 1896.25
   770.6 1902.51   782.6  1907.3   798.6 1909.16   814.7 1915.77     887 1937.16
#Mann= 5 ,-1,0
       0      .1       0  450.24    .045       0  564.17     .06       0
  637.85     .05       0  737.85      .1       0
Bank Sta=450.24,564.17
XS Rating Curve= 0 ,0
Exp/Cntr(USF)=0,0
Exp/Cntr=0.3,0.1

Type RM Length L Ch R = 1 ,38678   ,635.6,635.6,635.6
XS GIS Cut Line= 2
2229371.06745106689208.6317378292229641.68543374689882.046345055
#Sta/Elev= 30
       0 1928.99    86.8 1884.39   112.7 1872.91   133.5 1865.39   160.1 1861.31
   164.3 1858.61  174.911847.041   182.7  1844.8   228.8 1844.64   268.8 1844.72
  296.421847.042   348.8 1850.35   384.3 1848.01   413.3 1848.46     436 1854.49
   457.5 1853.05   479.1 1854.14   490.2 1858.33   500.7 1864.43     521 1866.58
   526.5 1868.77   548.1 1887.66     564 1889.76   573.9 1896.71   608.4 1907.63
   621.4 1909.97     686 1931.02     699 1932.42   707.6 1936.68   725.8 1941.69
#Mann= 5 ,-1,0
       0      .1       0  174.91    .045       0  296.42      .1       0
     510     .06       0     620      .1       0
Bank Sta=174.91,296.42
XS Rating Curve= 0 ,0
Exp/Cntr(USF)=0,0
Exp/Cntr=0.3,0.1

Type RM Length L Ch R = 1 ,38043   ,628,628,628
XS GIS Cut Line= 2
2228753.44326701 689428.375204382229098.14020908690108.309269387
#Sta/Elev= 30
       0 1934.46    11.6  1931.5    41.3 1929.78    68.1 1916.94   109.8 1899.95
   153.4 1880.61   171.3 1869.64   189.3 1864.85  225.721845.883   234.1 1842.59
   238.6 1841.87   274.5 1841.73   341.7 1841.98  349.441845.884   359.7 1848.02
   392.5 1849.09   413.5 1848.76   428.2 1847.03   444.9 1846.44   449.4 1847.09
   462.8  1855.3   476.3 1861.06   507.7 1862.78   547.2 1863.24   556.2 1866.74
   606.8 1877.15   654.4 1889.57   691.5 1900.48   722.8 1907.28   762.3 1920.26
#Mann= 5 ,-1,0
       0      .1       0  225.72    .045       0  349.44      .1       0
     510     .06       0     620      .1       0
Bank Sta=225.72,349.44
XS Rating Curve= 0 ,0
Exp/Cntr(USF)=0,0
Exp/Cntr=0.3,0.1

Type RM Length L Ch R = 1 ,37415   ,591.9,591.9,591.9
XS GIS Cut Line= 2
2228189.49456042689707.0914218412228551.49582201690369.796165049
#Sta/Elev= 30
       0 1949.74    34.3 1932.28    52.5 1924.52    66.2 1915.75    75.3 1913.14
    94.9 1911.07   120.9 1895.86   165.6 1876.22   175.6 1869.08   184.7 1867.39
   207.5 1867.24   216.6  1864.2   239.4 1860.96   243.9 1858.22   253.1 1849.81
  260.421845.311   266.7 1842.29   298.3 1840.97   371.6    1841  381.581845.312
   404.4 1853.55   412.6 1854.97   453.6 1855.79   499.2 1860.99     537  1860.1
   547.9 1863.72   587.2 1869.41   622.2 1877.13   676.9 1894.95   755.1 1918.14
#Mann= 5 ,-1,0
       0      .1       0  260.42    .045       0  381.58      .1       0
     430     .06       0     640      .1       0
Bank Sta=260.42,381.58
XS Rating Curve= 0 ,0
Exp/Cntr(USF)=0,0
Exp/Cntr=0.3,0.1

Type RM Length L Ch R = 1 ,36823   ,548.9,548.9,548.9
XS GIS Cut Line= 3
2227765.80508195689834.9075003082227714.47466562690068.435582395
2228032.65594952690659.662955689
#Sta/Elev= 30
       0 1902.83    30.1 1895.36   104.7 1881.41   121.1 1873.57   153.9 1874.85
   178.4 1868.09     203 1864.31   339.9 1860.48   374.5 1861.68   388.6 1856.96
   394.5 1852.51  400.581844.962   409.2 1840.12     517 1839.92   521.5 1841.82
  524.08 1844.96   530.3 1849.43   544.3 1852.27   577.6 1850.25   598.8 1858.49
     617  1860.2   644.2 1858.85   653.3 1861.59   735.1 1870.08   771.4 1882.04
   810.9 1887.41   844.1 1896.06   889.5 1899.33   902.4 1897.74   910.5 1900.16
#Mann= 6 ,-1,0
       0      .1       0  400.58    .045       0  524.08      .1       0
   579.1     .06       0   699.1      .1       0   849.1     .05       0
Bank Sta=400.58,524.08
XS Rating Curve= 0 ,0
Exp/Cntr(USF)=0,0
Exp/Cntr=0.3,0.1

Type RM Length L Ch R = 1 ,36274   ,754.5,754.5,754.5
XS GIS Cut Line= 2
2227091.44936125690119.0399389252227545.26441222690853.689258902
#Sta/Elev= 30
       0 1878.98    16.6 1873.81     106 1854.98   153.2 1853.05   164.8 1854.42
   228.8 1854.81   326.9 1858.19   350.4 1856.01   378.31844.704   383.3 1841.54
   394.4 1839.45   449.2 1839.19   482.1 1839.54  494.161844.707   505.6 1853.39
   519.7 1859.37   600.8 1863.01   632.8 1862.96   637.2 1864.14   646.6 1870.06
   670.5 1872.38   684.3  1877.5   712.5 1876.83   726.6 1884.32   731.3 1885.53
   760.6 1889.79   795.5 1900.35   807.1 1901.59   823.4 1906.07   863.5 1913.74
#Mann= 5 ,-1,0
       0      .1       0   378.3    .045       0  494.16      .1       0
     610     .06       0     640      .1       0
Bank Sta=378.3,494.16
XS Rating Curve= 0 ,0
Exp/Cntr(USF)=0,0
Exp/Cntr=0.3,0.1

Type RM Length L Ch R = 1 ,35519   ,583.7,583.7,583.7
XS GIS Cut Line= 3
2226477.42604847 690607.401067412226953.24459605690998.391904501
2227413.19377082691111.154007785
#Sta/Elev= 30
       0 1903.26    31.6 1892.78    53.2 1884.01    86.4 1866.89      97 1863.14
   112.3 1852.79   119.7 1850.95   138.2 1850.01  146.05 1844.25   148.5 1842.02
   153.8  1840.2   226.2 1839.22   236.3 1840.54     259 1840.72   262.4 1841.52
  265.86 1844.25     278  1851.3   307.3 1852.66   319.4    1859   495.4 1858.16
   525.7 1859.88   538.3 1858.92   548.9 1861.84   565.9 1860.85   620.6 1864.44
   766.1 1877.64   878.6 1889.44   952.5 1901.56  1025.3 1910.88  1089.4 1921.58
#Mann= 4 ,-1,0
       0      .1       0  146.05    .045       0  265.86     .07       0
     320      .1       0
Bank Sta=146.05,265.86
XS Rating Curve= 0 ,0
Exp/Cntr(USF)=0,0
Exp/Cntr=0.3,0.1

Type RM Length L Ch R = 1 ,34936   ,811.6,811.6,811.6
XS GIS Cut Line= 3
2226288.86060166691261.0307891732227078.80831886691347.616008583
2227531.52824931691214.899885803
#Sta/Elev= 30
       0 1881.65    27.5 1879.91    83.8 1863.45   136.1 1855.61   160.3 1854.14
   176.4 1850.16   188.4 1844.87   208.6 1844.37   212.6 1843.09   220.6 1838.28
   224.7 1837.97   318.6 1838.18   329.3 1840.16  335.471843.169   349.4 1849.85
   358.5 1855.97   381.6 1857.61   389.6 1860.97   494.3 1856.39   554.6 1857.34
   612.4 1863.71   699.5 1867.06   817.1 1875.79   883.6 1885.12   933.7 1886.36
  1033.7 1899.38  1094.3 1904.89  1167.1 1919.21  1221.3 1934.22  1266.5 1943.02
#Mann= 5 ,-1,0
       0      .1       0      40     .06       0   212.6    .045       0
  335.47     .06       0     540      .1       0
#XS Ineff= 2 , 0
                          389.37         1872.06
Permanent Ineff=
       F       F
Bank Sta=212.6,335.47
XS Rating Curve= 0 ,0
Exp/Cntr(USF)=0,0
Exp/Cntr=0.3,0.1

Type RM Length L Ch R = 1 ,34124   ,631.8,631.8,631.8
XS GIS Cut Line= 2
2226207.45046147691998.4961916712227684.97284433692383.445400493
#Sta/Elev= 30
       0 1909.75    58.6 1899.75    87.6 1885.85   104.4 1869.07   124.8 1866.29
   152.41843.866   174.4 1836.76   281.8 1836.96  295.331843.865   327.3 1847.56
   339.7 1854.14     381 1856.17     410 1855.43   434.8 1846.32   455.4 1853.79
   476.1 1852.82   500.9 1846.46   517.6 1851.38     534 1848.14   575.3 1851.78
   620.8 1846.02   674.5  1846.6   703.4 1850.65     782 1846.28   881.2  1855.6
  1025.8 1860.94  1067.2 1858.85  1133.3 1869.05  1406.3  1889.2  1526.8 1915.93
#Mann= 5 ,-1,0
       0      .1       0     130     .06       0   152.4    .045       0
  295.33     .06       0     430      .1       0
#XS Ineff= 2 , 0
                          380.78         1864.85
Permanent Ineff=
       F       F
Bank Sta=152.4,295.33
XS Rating Curve= 0 ,0
Exp/Cntr(USF)=0,0
Exp/Cntr=0.3,0.1

Type RM Length L Ch R = 1 ,33492   ,713.4,713.4,713.4
XS GIS Cut Line= 4
 2226070.1481958691980.4648128692226029.17407345692228.524001464
2226123.34686556692646.415766461 2226101.7656007692773.941422446
#Sta/Elev= 30
       0 1909.73    41.3 1899.03   142.6 1875.44   195.3    1865   235.9  1861.2
     330 1857.72   383.3 1858.94   416.1 1858.28   436.6 1856.66   440.7 1854.93
     453 1845.72   469.4 1845.05  474.091843.691   481.7  1836.6   485.8 1835.88
   572.4 1835.92   580.1 1837.34     5931843.695   608.8  1847.5   621.1  1854.9
   625.2    1856   645.7 1856.22   649.8 1857.45   662.1 1858.13   669.4 1860.93
   679.4 1861.91     711 1871.33   723.2 1874.03   743.9 1880.13   809.1 1903.57
#Mann= 5 ,-1,0
       0      .1       0  471.42     .07       0  474.09    .045       0
     593     .06       0  769.79      .1       0
Bank Sta=474.09,593
XS Rating Curve= 0 ,0
Exp/Cntr(USF)=0,0
Exp/Cntr=0.3,0.1

Type RM Length L Ch R = 1 ,32779   ,433.4,433.4,433.4
XS GIS Cut Line= 2
2225706.76209965691849.9393946772225399.57085526692581.539198582
#Sta/Elev= 30
       0    1920    20.9 1913.74    47.2 1908.73    89.3  1898.5   116.3 1893.19
   185.7 1876.32   198.7 1874.98   216.1 1871.18   259.5 1864.65   285.5 1861.88
   294.2 1860.02   337.6 1855.84   415.7 1843.95   441.4 1842.83   453.6  1840.1
   461.3  1837.2     475 1834.15   487.3 1833.66   550.1 1833.95   563.2 1836.71
  569.151840.237   580.5 1846.91   595.6 1850.44   623.9 1854.76   645.6  1855.7
   661.4 1857.42   732.3  1867.6     750 1871.61   775.7 1880.13   793.5 1882.17
#Mann= 5 ,-1,0
       0      .1       0     320     .06       0   453.6    .045       0
  569.15      .1       0     750     .06       0
Bank Sta=453.6,569.15
XS Rating Curve= 0 ,0
Exp/Cntr(USF)=0,0
Exp/Cntr=0.3,0.1

Type RM Length L Ch R = 1 ,32345   ,504.4,504.4,504.4
XS GIS Cut Line= 2
2225309.08972194691696.4761488292225053.77779171 692432.14842801
#Sta/Elev= 30
       0 1919.46      15 1917.28    47.3 1907.03   110.8 1891.45     187  1875.3
   243.3 1867.05   292.9 1861.67   326.8 1859.87     331 1858.85   339.5 1851.24
   343.7 1849.23   360.6 1848.21   364.9 1847.15   377.6 1840.86     386 1839.89
   398.7 1834.46     403 1834.06   466.4 1833.66   491.6 1834.33   496.1 1836.05
   500.4 1839.92   504.6 1843.97   513.1  1846.4     530 1845.86     585 1853.29
   606.2 1855.05   633.1 1855.55   665.5 1860.57   690.9 1866.61   778.7 1893.45
#Mann= 4 ,-1,0
       0      .1       0     260     .06       0     386    .045       0
   500.4      .1       0
Bank Sta=386,500.4
XS Rating Curve= 0 ,0
Exp/Cntr(USF)=0,0
Exp/Cntr=0.3,0.1

Type RM Length L Ch R = 1 ,31841   ,503.2,503.2,503.2
XS GIS Cut Line= 2
2224875.55737008691504.5706621032224585.19126107692299.153595548
#Sta/Elev= 30
       0 1949.32    51.8    1925   119.9 1907.97   158.2 1895.14     188 1886.74
   213.6 1877.53   247.7 1874.75   274.5 1868.65   345.6 1857.82   409.5  1855.7
   433.5 1856.06   443.6 1851.29   464.4 1851.12   469.1 1849.74   477.6 1845.13
   483.4 1839.67   486.1  1836.4   489.7 1834.12   494.7 1833.43   579.8 1833.31
   588.4 1834.18   596.41839.662   605.4 1841.04   622.4 1849.15   635.2 1852.06
   660.7 1855.79   673.5 1855.49   699.1 1861.07   818.3 1896.25     846 1903.16
#Mann= 4 ,-1,0
       0      .1       0     370     .06       0   483.4    .045       0
   596.4      .1       0
Bank Sta=483.4,596.4
XS Rating Curve= 0 ,0
Exp/Cntr(USF)=0,0
Exp/Cntr=0.3,0.1

Type RM Length L Ch R = 1 ,31338   ,761.9,761.9,761.9
XS GIS Cut Line= 4
2224519.12098514691232.7052649022224336.48599968691435.960354381
2224158.40708067692057.2722123972224195.82316923 692240.52084286
#Sta/Elev= 30
       0 1961.64    30.7 1957.72    54.4 1950.61    76.1 1942.52   132.7 1916.05
   156.6  1907.3   291.2 1874.99   378.5 1863.23     520 1855.91     570 1855.25
   597.9 1856.82   607.6 1852.03   632.4 1851.39   644.9 1842.65   653.7 1840.66
   662.6 1834.14   678.1 1833.22   743.4 1833.53   765.5 1836.03   772.5 1840.66
     778 1842.14   819.6 1842.72   832.1 1840.59   836.3 1841.66   844.6 1848.12
   861.2 1855.11   915.3 1858.24   948.1 1863.88  1030.1 1873.69  1106.6  1887.2
#Mann= 4 ,-1,0
       0      .1       0  493.25     .06       0   653.7    .045       0
   772.5      .1       0
Bank Sta=653.7,772.5
XS Rating Curve= 0 ,0
Exp/Cntr(USF)=0,0
Exp/Cntr=0.3,0.1

Type RM Length L Ch R = 1 ,30576   ,668.1,668.1,668.1
XS GIS Cut Line= 4
2223495.95165029690997.5980265162223605.08434569691164.521015617
2223452.48954365691929.6749515262223755.78595837692297.515920726
#Sta/Elev= 30
       0 1977.49    43.2 1955.57    99.9 1936.37   118.3 1927.21   128.5 1926.31
   166.8 1905.05   187.7 1886.06   208.3 1883.47   228.7 1871.33   261.3 1862.15
   281.7 1848.53   318.4 1846.46   338.8 1851.17   563.1 1855.57     608 1853.83
   620.2 1846.58   632.6 1842.78   665.1 1842.22   742.6 1837.92   768.7 1842.18
   828.2 1854.61   893.5 1855.17   991.7 1860.99  1113.8 1863.46  1209.2 1862.13
    1303 1867.55    1325 1861.68  1345.6 1869.92  1419.5 1875.47  1456.4 1882.74
#Mann= 10 ,-1,0
       0      .1       0     140     .06       0     190     .08       0
  399.43      .1       0  599.43     .08       0   665.1    .045       0
   768.7      .1       0  799.43     .05       0 1169.65     .07       0
 1329.65     .05       0
Bank Sta=665.1,768.7
XS Rating Curve= 0 ,0
Exp/Cntr(USF)=0,0
Exp/Cntr=0.3,0.1

Type RM Length L Ch R = 1 ,29908   ,739.7,739.7,739.7
XS GIS Cut Line= 3
2222847.14983254691374.4463501112223081.90216729691953.654134703
 2223754.3703708692312.052905947
#Sta/Elev= 30
       0 1926.85    13.4 1925.95    20.2  1921.3    41.8 1902.15      72 1870.55
    93.6 1844.03  101.741838.269   110.8 1833.79   132.4 1832.78   190.2 1833.31
   192.9 1833.74  198.231838.271   201.5 1841.02   214.4 1844.63   261.9 1851.26
   300.9 1854.35   466.6 1854.41   520.9 1851.19   681.9 1861.07   871.7 1856.27
  1035.5  1854.4  1117.1 1855.91  1199.9 1861.02  1239.5 1865.17  1259.1 1861.15
  1262.1 1861.72  1271.2 1867.63  1316.5 1871.07  1356.6 1878.01    1387 1885.29
#Mann= 7 ,-1,0
       0     .06       0      90      .1       0  101.74    .045       0
  198.23      .1       0     300     .05       0 1184.97     .07       0
 1234.97     .05       0
#XS Ineff= 2 , 0
                          372.75         1864.47
Permanent Ineff=
       F       F
Bank Sta=101.74,198.23
XS Rating Curve= 0 ,0
Exp/Cntr(USF)=0,0
Exp/Cntr=0.3,0.1
