HEC-RAS study MIDFKRIV.prj: MIDFKRIV

--- MIDFKRIV.g01 (geometry) --- (continued)

Type RM Length L Ch R = 1 ,29168   ,551.3,551.3,551.3
XS GIS Cut Line= 3
2222317.13164172691430.3870034612222328.48342563691957.031929642
2223734.94913055692325.788416989
#Sta/Elev= 30
       0 1956.37    70.8 1924.35   114.8 1907.89   126.8 1899.27   146.8 1899.17
   158.8 1893.71   238.8 1868.13   295.5 1854.07   366.9 1849.78   414.9 1844.81
   426.9 1841.77  432.361837.405   446.9 1831.57     515 1831.54  532.991837.409
   574.7 1849.55   588.5 1850.57     605 1854.47     634 1855.53     940 1854.55
  1073.8 1851.08  1456.9 1851.66  1655.4 1850.92  1697.5 1849.18  1787.7 1855.76
  1845.6 1862.11  1866.3 1859.92  1879.7 1865.01  1925.6 1868.66  1980.8 1881.13
#Mann= 6 ,-1,0
       0      .1       0     120     .06       0     220      .1       0
  432.36    .045       0  532.99      .1       0  596.77     .05       0
#XS Ineff= 2 , 0
                          763.14         1864.67
Permanent Ineff=
       F       F
Bank Sta=432.36,532.99
XS Rating Curve= 0 ,0
Exp/Cntr(USF)=0,0
Exp/Cntr=0.3,0.1

Type RM Length L Ch R = 1 ,28617   ,533.6,533.6,533.6
XS GIS Cut Line= 3
2221832.72706839692322.8437539852222136.50921441692123.199441189
2223738.77446783692338.366475247
#Sta/Elev= 30
       0 1932.11    38.4 1916.28    44.1 1912.74      54 1902.81    71.1    1902
    90.3 1889.59   109.4 1866.86   141.4 1836.86   152.5 1831.79   159.8 1830.97
   238.7 1830.99   249.2 1833.54  254.841836.799   267.4  1843.7   309.9 1842.18
   324.8 1844.93     344 1852.36   358.3 1854.31   415.6 1852.77   665.9 1852.97
   916.5 1855.39    1134 1851.61  1412.5 1852.28  1738.4 1848.97  1836.3 1860.72
  1856.5 1859.05  1868.6 1863.39    1913 1866.51  1945.3 1871.79  1980.2 1881.01
#Mann= 4 ,-1,0
       0      .1       0   141.4    .045       0  254.84      .1       0
  423.51     .05       0
#XS Ineff= 2 , 0
                          359.44         1862.96
Permanent Ineff=
       F       F
Bank Sta=141.4,254.84
XS Rating Curve= 0 ,0
Exp/Cntr(USF)=0,0
Exp/Cntr=0.3,0.1

Type RM Length L Ch R = 1 ,28083   ,783.1,783.1,783.1
XS GIS Cut Line= 3
2222308.28242617692649.7319632512222520.31689104692318.899603035
 2223763.3391532692374.056978048
#Sta/Elev= 30
       0 1919.42    32.2 1896.67    71.9 1873.38    81.4 1864.27   101.7 1861.91
   121.9 1852.85   162.5 1851.53   208.8  1846.3  232.231836.959   247.7  1830.8
   274.1 1830.72   342.7 1830.93   347.5 1832.18  355.861836.958   361.7 1841.45
     376 1849.18   392.9 1853.98     625 1854.44   789.2 1851.67   881.3 1853.74
   945.3 1852.53  1021.4 1854.33  1197.6 1853.92  1293.7 1852.95  1313.7 1849.45
  1328.9 1848.83  1405.8 1850.28  1545.1 1865.96    1594 1873.97  1637.2 1884.14
#Mann= 4 ,-1,0
       0      .1       0  232.23    .045       0  355.86      .1       0
  462.95     .05       0
#XS Ineff= 2 , 0
                          640.02          1859.2
Permanent Ineff=
       F       F
Bank Sta=232.23,355.86
XS Rating Curve= 0 ,0
Exp/Cntr(USF)=0,0
Exp/Cntr=0.3,0.1

Type RM Length L Ch R = 1 ,27300   ,849.6,849.6,849.6
XS GIS Cut Line= 3
 2222905.9900221693130.2265643772223343.19265774692504.949432625
2223829.48468336692483.918180626
#Sta/Elev= 30
       0 1904.59      55 1885.69   122.5 1857.91   131.6 1851.67   143.1 1851.33
   157.4 1846.69   186.2 1843.82   206.2 1836.29   222.6 1835.75   235.6 1830.53
   338.4 1830.53   342.9 1831.13  347.631835.839   352.8 1840.05   362.5 1843.32
   372.2 1849.85     382 1852.84   588.3  1846.3   665.1 1847.64   723.6 1851.61
     800 1853.68   822.8 1853.37     860 1849.37   908.1 1850.43   988.2 1847.94
  1012.2 1855.84  1036.2 1853.38  1084.2 1859.55  1170.2  1878.1  1249.7 1898.42
#Mann= 4 ,-1,0
       0      .1       0   222.6    .045       0  347.63      .1       0
     480     .05       0
#XS Ineff= 2 , 0
                          384.62         1857.64
Permanent Ineff=
       F       F
Bank Sta=222.6,347.63
XS Rating Curve= 0 ,0
Exp/Cntr(USF)=0,0
Exp/Cntr=0.3,0.1

Type RM Length L Ch R = 1 ,26450   ,865.3,865.3,865.3
XS GIS Cut Line= 2
2223285.19291221693490.5080106782224048.61152636693041.084244031
#Sta/Elev= 30
       0 1879.84      22  1873.3    70.3 1863.81   117.1 1855.98   155.1 1852.05
   210.6 1850.03   319.1 1848.83   407.3 1850.24   505.7  1849.8   551.2 1847.42
   562.4 1843.97   569.7 1840.26     579  1838.3  584.261836.013     593 1830.52
   597.6 1830.22   685.8 1830.22  694.99 1836.01   704.4 1842.87     709 1848.06
     716 1853.57   736.8  1858.1   741.5 1861.77   764.7 1886.77   792.5  1900.9
   820.4 1918.28   852.9 1933.67   876.1 1934.46   880.7 1937.62   885.9 1943.54
#Mann= 4 ,-1,0
       0      .1       0  584.26    .045       0  694.99      .1       0
     790     .06       0
Bank Sta=584.26,694.99
XS Rating Curve= 0 ,0
Exp/Cntr(USF)=0,0
Exp/Cntr=0.3,0.1

Type RM Length L Ch R = 1 ,25585   ,277.4,277.4,277.4
XS GIS Cut Line= 2
2223362.83099682694025.4354663892224288.89497444693826.348990964
#Sta/Elev= 30
       0 1911.32    42.3 1894.93    95.6 1868.04   136.4 1854.43   144.6 1850.05
   186.6 1847.92  210.051835.423   218.2 1830.08   222.3 1829.78   320.5 1829.89
  326.721835.428   332.8 1839.93   343.8  1840.8   357.3 1846.01   377.8 1849.27
   492.3 1847.97   541.4 1849.23     611 1855.86   641.2 1856.71   668.3 1862.07
   692.8 1862.53   741.9 1867.82     791  1877.2   815.6 1880.15   831.9 1890.61
   856.5 1891.02   868.7 1899.39   907.2  1917.7   930.1 1926.27   947.2 1930.36
#Mann= 7 ,-1,0
       0      .1       0  210.05    .045       0  326.72      .1       0
     420     .05       0     520      .1       0     820     .06       0
     920      .1       0
Bank Sta=210.05,326.72
XS Rating Curve= 0 ,0
Exp/Cntr(USF)=0,0
Exp/Cntr=0.3,0.1

Type RM Length L Ch R = 1 ,25308   ,652.6,652.6,652.6
XS GIS Cut Line= 2
2223398.63855341694375.2140728892224204.84756504693975.413702363
#Sta/Elev= 30
       0 1922.57      24 1913.86    82.1 1897.57   148.9 1867.25   181.7 1855.49
   193.7 1848.03   211.6 1846.79   232.5 1832.62   242.8 1829.66   342.9 1829.71
   348.9 1830.73   353.4 1833.83   358.9 1837.42   382.7 1841.28   396.6 1847.83
   414.6 1850.22   537.5 1843.39   550.9 1839.91   573.2 1844.81   604.5 1847.21
   640.2 1848.25   671.4 1845.96   688.8 1850.72   706.9 1850.98   756.3 1856.79
   769.7  1862.9   796.5 1866.68   872.4  1883.9   890.2 1891.74   899.9  1892.2
#Mann= 4 ,-1,0
       0      .1       0   232.5    .045       0   353.4      .1       0
     860     .06       0
Bank Sta=232.5,353.4
XS Rating Curve= 0 ,0
Exp/Cntr(USF)=0,0
Exp/Cntr=0.3,0.1

Type RM Length L Ch R = 1 ,24655   ,506,506,506
XS GIS Cut Line= 2
2223505.00994551694641.8707480582224431.41500596694568.179445277
#Sta/Elev= 30
       0 1911.24   103.5 1874.79   139.6 1866.18   151.6 1864.61   175.7 1857.56
     256 1852.69   292.1 1848.29   356.3 1849.47   548.9 1846.47     589 1841.86
   605.1 1837.28  609.181834.781   617.1 1829.88   621.1 1829.34   721.4 1829.34
   725.4 1829.75  728.541834.778   733.5 1841.31   745.5 1852.56   769.6 1853.95
   777.6 1859.53   785.6 1867.43   797.7 1875.11   813.7 1877.44   821.8 1884.95
   829.8 1887.28   849.8    1898   861.9 1907.85     890 1909.37   929.3 1921.62
#Mann= 5 ,-1,0
       0      .1       0  609.18    .045       0  728.54      .1       0
     760     .06       0     860      .1       0
Bank Sta=609.18,728.54
XS Rating Curve= 0 ,0
Exp/Cntr(USF)=0,0
Exp/Cntr=0.3,0.1

Type RM Length L Ch R = 1 ,24149   ,506.1,506.1,506.1
XS GIS Cut Line= 2
2223579.39326685695136.2635087932224484.03337386695073.242504728
#Sta/Elev= 30
       0 1924.67    64.9  1905.8      97 1899.17   189.2 1862.76   217.3 1854.53
   245.4 1849.42   316.5 1845.89   465.9 1848.26   477.9 1839.57     486  1836.6
     510 1835.99   526.1 1838.55   534.1 1837.74  539.231834.527   546.1 1829.69
   554.1 1828.28   654.4 1828.31  662.171834.528   686.4 1850.69   702.5 1855.61
   710.5 1860.54   718.5 1868.53   726.5 1879.71   734.5 1884.95   754.6 1886.72
   766.6 1893.86   822.8  1912.7   866.9 1920.84   890.9 1920.83   906.8 1930.72
#Mann= 5 ,-1,0
       0      .1       0  539.23    .045       0  662.17      .1       0
     790     .06       0     890      .1       0
Bank Sta=539.23,662.17
XS Rating Curve= 0 ,0
Exp/Cntr(USF)=0,0
Exp/Cntr=0.3,0.1

Type RM Length L Ch R = 1 ,23643   ,442.9,442.9,442.9
XS GIS Cut Line= 3
 2223536.9925379695505.7523419822223718.15320897695591.292560311
2224503.39204698695538.401734383
#Sta/Elev= 30
       0 1937.94    47.8  1919.5    69.9 1912.67   149.5 1900.61   226.4 1880.05
   286.6  1852.5   302.6 1842.35   318.6 1842.75   338.7 1840.42   370.7 1846.32
   390.8 1846.72   394.8 1846.08   406.8 1836.97  428.251834.323   438.9 1829.03
   446.9 1827.89   543.1 1827.94   551.2  1830.1   556.91834.321   579.2 1844.52
   587.1 1846.43   627.3 1846.27   688.8 1852.27   715.5 1852.98   779.7 1860.31
   787.7 1862.82   862.2 1872.94     904 1876.62     928 1884.01   987.4 1908.36
#Mann= 6 ,-1,0
       0      .1       0  428.25    .045       0   556.9      .1       0
  650.34     .08       0  750.34      .1       0  950.34     .06       0
Bank Sta=428.25,556.9
XS Rating Curve= 0 ,0
Exp/Cntr(USF)=0,0
Exp/Cntr=0.3,0.1

Type RM Length L Ch R = 1 ,23200   ,566.2,566.2,566.2
XS GIS Cut Line= 4
 2223728.7248893696285.8803833712223868.52719896696089.406402163
2224332.18033478695823.1191282172224524.12298885695775.164117856
#Sta/Elev= 30
       0 1906.49    64.7 1899.84   109.1 1892.21     137 1885.53   192.5 1868.62
   212.9 1863.59   226.7 1861.46   236.5 1856.63   259.2 1856.98   360.7 1844.88
     370 1840.89  378.751834.097   383.7 1831.03     393 1827.57   397.6 1827.34
   472.5 1827.45   478.4 1828.83  488.641834.098   494.4 1835.82   504.7 1836.01
   517.5 1839.43   674.3  1848.4   718.6 1849.76   788.2 1856.86   836.8 1864.51
   870.6 1870.92   882.8 1874.31   891.3 1874.94   944.9 1891.39   973.7 1901.47
#Mann= 5 ,-1,0
       0      .1       0  378.75    .045       0  488.64      .1       0
  581.14     .05       0  701.14      .1       0
Bank Sta=378.75,488.64
XS Rating Curve= 0 ,0
Exp/Cntr(USF)=0,0
Exp/Cntr=0.3,0.1

Type RM Length L Ch R = 1 ,22634   ,507.9,507.9,507.9
XS GIS Cut Line= 2
 2224250.9953978696675.1566325152224631.45659488695953.375291843
#Sta/Elev= 30
       0 1950.34    56.5 1927.46    70.1 1921.29    76.4 1917.06    88.1 1915.23
    97.1 1909.56   142.4 1887.63   153.3 1879.56   169.5 1878.18   174.1 1876.38
   183.1 1869.09   205.7 1855.83   221.4 1841.08   231.4 1833.81   239.2 1828.06
   246.4 1827.12   327.8 1827.18   337.91833.813   341.4    1835   366.5 1836.47
   382.1 1842.38   400.1 1842.83   422.8 1845.94   567.4 1846.46   591.6 1847.36
   635.3 1851.68   671.5 1857.26   698.6 1864.11   766.3  1878.2   815.9 1894.94
#Mann= 5 ,-1,0
       0      .1       0   231.4    .045       0   337.9      .1       0
     460     .05       0     680      .1       0
Bank Sta=231.4,337.9
XS Rating Curve= 0 ,0
Exp/Cntr(USF)=0,0
Exp/Cntr=0.3,0.1

Type RM Length L Ch R = 1 ,22126   ,527.6,527.6,527.6
XS GIS Cut Line= 2
2224909.07120866696717.4085508442224850.42249991695995.717431786
#Sta/Elev= 30
       0 1892.97     8.3  1892.5    24.3 1886.03    76.5 1873.14   136.7 1864.22
   169.6 1857.82   196.9 1855.16     222 1848.42     237 1845.51   257.1 1838.13
   260.9 1836.01  262.971833.572   265.1  1830.9   269.1 1828.09   277.1    1827
   364.8  1827.2  378.181833.577   381.5 1835.91   393.5 1834.87   405.5 1837.99
   441.7 1844.34   489.8 1845.05   521.9 1846.97   562.1  1853.1   590.2 1860.72
   610.2 1862.62   630.3 1869.41   670.4 1879.02     710 1890.34   724.1 1895.66
#Mann= 6 ,-1,0
       0      .1       0  262.97    .045       0  378.18      .1       0
     450     .05       0     650     .06       0     710      .1       0
Bank Sta=262.97,378.18
XS Rating Curve= 0 ,0
Exp/Cntr(USF)=0,0
Exp/Cntr=0.3,0.1

Type RM Length L Ch R = 1 ,21599   ,500.2,500.2,500.2
XS GIS Cut Line= 3
2225320.97309492696824.207470484  2225308.044874696618.848158598
2225591.68925696695934.223324535
#Sta/Elev= 30
       0 1903.74    71.5 1876.64    97.9 1870.18   155.3 1862.61   175.4 1860.92
   268.4  1847.4   285.5 1846.39   367.8 1846.85   393.8 1838.76   398.1 1836.69
  401.99 1833.38   406.7 1829.39   411.1 1827.34   415.3 1826.97   519.3 1826.97
     528 1828.81  540.121833.382   563.4  1839.5   575.6 1840.35   592.9 1846.41
   614.6 1846.53     645 1850.67   670.9 1851.22   679.5 1853.61   770.4 1863.53
   848.4 1879.56     896 1893.81   917.4 1902.03   927.2 1907.14   946.8 1910.62
#Mann= 5 ,-1,0
       0      .1       0  401.99    .045       0  540.12      .1       0
  565.77     .06       0  695.77      .1       0
Bank Sta=401.99,540.12
XS Rating Curve= 0 ,0
Exp/Cntr(USF)=0,0
Exp/Cntr=0.3,0.1

Type RM Length L Ch R = 1 ,21098   ,540.2,540.2,540.2
XS GIS Cut Line= 2
2225664.04313321 696990.051350982226064.02596058696102.608245154
#Sta/Elev= 30
       0 1906.45    27.3 1902.93    43.1 1899.04   128.2 1871.41   167.7 1864.38
   185.3  1863.3   197.3 1859.18   233.6 1852.94   286.1 1847.19   325.6 1845.13
   369.7 1843.92   430.2 1845.28   452.9 1842.75   472.6 1836.69  497.491833.114
   509.9 1828.39   518.7 1826.97     602 1826.99   606.4 1828.99  610.331833.116
   626.8 1846.42   632.5 1848.46   667.9 1849.73   707.3 1854.59   795.1 1869.01
   830.2 1876.08   847.7 1877.45   869.7 1881.32   925.1 1893.77   973.4 1911.96
#Mann= 5 ,-1,0
       0      .1       0  497.49    .045       0  610.33      .1       0
     660     .07       0     680      .1       0
Bank Sta=497.49,610.33
XS Rating Curve= 0 ,0
Exp/Cntr(USF)=0,0
Exp/Cntr=0.3,0.1

Type RM Length L Ch R = 1 ,20558   ,363.4,363.4,363.4
XS GIS Cut Line= 3
2226095.10681935697179.3082981682226511.03679395696455.943002772
2226653.75965994696410.584280792
#Sta/Elev= 30
       0 1887.05    52.1 1876.15   168.6 1858.36   270.1 1848.94   297.8 1847.89
  332.891832.734     348 1827.92   376.2 1826.84   436.2 1826.85   444.7 1829.17
  449.371832.735   465.2 1841.92   477.7 1843.37   500.4 1843.38   547.8 1837.89
   573.6 1839.47     612 1838.93   634.6 1846.59   649.8 1848.34   662.3 1853.67
   676.1 1852.87     713 1855.86   731.5 1865.83   749.9  1867.3   775.8 1874.99
   822.6 1877.28     833 1880.64   856.6 1896.03   890.2 1911.04   984.2 1946.11
#Mann= 5 ,-1,0
       0      .1       0  332.89    .045       0  449.37      .1       0
     670     .06       0     820      .1       0
Bank Sta=332.89,449.37
XS Rating Curve= 0 ,0
Exp/Cntr(USF)=0,0
Exp/Cntr=0.3,0.1

Type RM Length L Ch R = 1 ,20195   ,243.2,243.2,243.2
XS GIS Cut Line= 3
2226164.30452741697331.8036755682226710.27984332696874.147896051
2226798.59937972696764.417562951
#Sta/Elev= 30
       0 1898.67    30.2 1893.26    98.3 1877.72   161.6 1861.08   183.5  1860.4
   198.2  1857.2   239.9 1853.39   380.8 1846.26   504.3 1846.34   521.8 1843.69
   532.2 1838.98   541.2  1837.5  549.54 1832.21   553.1 1828.74   558.3 1826.63
   657.9 1826.62   664.1 1827.25   673.1 1832.17   691.7 1843.87   718.8 1847.17
   734.2 1854.16   747.3 1856.07   754.7 1862.79   759.9 1865.71   782.7 1867.24
   791.3 1874.15   805.5 1890.36     843 1917.96   848.2 1920.73   853.3 1921.65
#Mann= 3 ,0,0
       0      .1       0  549.54    .045       0   673.1      .1       0
Bank Sta=549.54,673.1
XS Rating Curve= 0 ,0
Exp/Cntr(USF)=0,0
Exp/Cntr=0.3,0.1

Type RM Length L Ch R = 1 ,19951   ,502.8,502.8,502.8
XS GIS Cut Line= 2
2226284.12181712697509.5739243162227018.67217574696950.788235178
#Sta/Elev= 30
       0 1899.25    80.2 1877.08     191 1854.75   391.4 1844.41   459.9  1845.9
   502.7 1845.35     516 1844.01   532.8 1840.15   547.9 1835.19  552.021832.407
   562.6 1827.49     568  1826.5     674 1826.52   678.6 1827.53  684.771832.409
   713.9 1853.11   718.8 1855.09     734  1857.6   753.9 1874.05   759.6 1876.02
   779.1 1876.31   784.1 1879.07     791  1885.3   799.2 1898.28   802.4 1901.75
   829.3  1922.7   842.4 1926.91   850.9 1932.85     886 1952.33   922.9 1976.38
#Mann= 4 ,-1,0
       0      .1       0  552.02    .045       0  684.77     .06       0
     910      .1       0
Bank Sta=552.02,684.77
XS Rating Curve= 0 ,0
Exp/Cntr(USF)=0,0
Exp/Cntr=0.3,0.1

Type RM Length L Ch R = 1 ,19449   ,512.5,512.5,512.5
XS GIS Cut Line= 2
2226588.27042826 697798.980648632227268.63828025697443.272673487
#Sta/Elev= 30
       0 1878.01    22.5 1874.83    58.6 1866.67    85.7 1862.38    94.7 1858.84
   110.9  1859.9   121.8 1855.49   135.3 1853.26   259.1 1844.09   356.5 1844.04
   377.7 1841.58   401.4 1834.78   418.3 1834.36  424.511832.098   433.2 1826.79
   437.7 1826.47   531.8 1826.49     537 1828.01  542.411832.097   573.3 1850.34
     591 1855.13   618.3  1878.8   625.5 1880.51   645.3 1880.97   649.9 1883.94
     660 1894.32   697.8 1920.51     704 1922.65   717.6 1932.21   767.7 1957.71
#Mann= 5 ,-1,0
       0      .1       0  424.51    .045       0  542.41      .1       0
     600     .06       0     710      .1       0
Bank Sta=424.51,542.41
XS Rating Curve= 0 ,0
Exp/Cntr(USF)=0,0
Exp/Cntr=0.3,0.1

Type RM Length L Ch R = 1 ,18936   ,449.8,449.8,449.8
XS GIS Cut Line= 2
2226830.60143365698218.6890746242227508.37555322697915.836469329
#Sta/Elev= 30
       0 1906.18    80.6 1879.44    90.1 1874.59   106.9 1873.17   124.4 1867.15
   150.8 1862.36   174.9 1856.12   219.4 1848.13   247.1  1844.3   290.9 1842.21
   305.1 1837.63   317.2 1837.41   325.9 1834.25  344.381831.792   356.5 1826.65
     361 1826.44   474.9 1826.44   479.3 1827.88  484.931831.794   495.9 1838.87
   514.1 1846.58   536.2 1846.93     545 1851.05   562.5  1854.2   571.3 1858.39
     611 1858.46   621.4 1864.47   663.3 1879.46   724.6  1905.8   742.4 1914.48
#Mann= 5 ,-1,0
       0      .1       0  344.38    .045       0  484.93      .1       0
     530     .06       0     670      .1       0
Bank Sta=344.38,484.93
XS Rating Curve= 0 ,0
Exp/Cntr(USF)=0,0
Exp/Cntr=0.3,0.1

Type RM Length L Ch R = 1 ,18486   ,423.9,423.9,423.9
XS GIS Cut Line= 3
2227036.06300225698539.8139298912227569.92030682698424.902434246
2227731.33243249698286.473826132
#Sta/Elev= 30
       0 1866.27    24.7 1858.36      41 1856.88    57.4 1851.09   110.6 1842.87
   163.8 1839.99     172 1835.48   192.4 1833.84   204.7 1839.21   217.8 1839.95
   225.2  1839.1   245.6 1832.05  266.391831.413   274.3 1827.53   282.4 1826.41
   376.5  1826.5  388.751831.411   421.6 1847.09   478.8 1846.71   493.9 1847.61
   519.7 1852.68   540.2 1853.17   591.2 1864.84   607.1 1866.54   622.8 1871.48
   638.6 1873.18   668.5 1879.57   692.2 1887.13   748.4 1914.21   758.7 1917.25
#Mann= 5 ,-1,0
       0      .1       0  266.39    .045       0  388.75      .1       0
     390     .06       0     490      .1       0
Bank Sta=266.39,388.75
XS Rating Curve= 0 ,0
Exp/Cntr(USF)=0,0
Exp/Cntr=0.3,0.1

Type RM Length L Ch R = 1 ,18062   ,438.6,438.6,438.6
XS GIS Cut Line= 3
2227120.38975485698978.7948724962227869.10189108698692.756103921
2227957.90196696698518.743571699
#Sta/Elev= 30
       0 1896.37    42.6 1875.03      60 1869.68    76.8 1855.42   102.5 1853.76
   121.9 1845.32   136.8 1844.14   153.9 1835.67   168.4 1833.08  173.66 1830.86
   179.6 1826.83     187 1826.32   276.8 1826.39  289.981830.859   308.1 1835.18
   320.9  1842.7   346.6 1843.58   359.5 1845.94   376.6  1844.7   441.6 1845.39
   513.6 1844.19   612.1 1846.46   659.2 1845.93   766.4 1856.34   803.5  1860.8
   832.5 1866.09   848.1 1865.85   913.3 1877.77   958.5 1889.56   996.9  1893.2
#Mann= 5 ,-1,0
       0      .1       0  173.66    .045       0  289.98      .1       0
     320     .06       0     420      .1       0
Bank Sta=173.66,289.98
XS Rating Curve= 0 ,0
Exp/Cntr(USF)=0,0
Exp/Cntr=0.3,0.1

Type RM Length L Ch R = 1 ,17624   ,403.1,403.1,403.1
XS GIS Cut Line= 3
2227263.96096972 699346.152556252228201.17778564699168.940405566
2228327.53158799699358.655359367
#Sta/Elev= 30
       0 1912.05    49.1 1876.22    69.4 1853.65    93.8 1836.58   150.8 1833.58
   162.31830.337   167.1 1826.52   171.2 1825.91   301.5 1825.94  312.851830.278
   382.9 1830.04   403.2 1834.36   427.7 1835.92   452.1 1840.25     505 1838.44
   637.8 1841.62   663.8 1843.85   684.1 1842.05   785.9 1843.62   834.7 1850.76
   895.8 1848.83   920.2 1846.14   953.8 1847.79  1088.7 1875.05  1110.8 1882.08
  1122.3 1887.89  1132.4 1889.22  1146.3 1897.23  1165.6 1904.22  1181.8 1912.79
#Mann= 8 ,-1,0
       0      .1       0   162.3    .045       0  312.85      .1       0
     350     .05       0     450     .08       0     550     .05       0
     860     .06       0  953.82      .1       0
Bank Sta=162.3,312.85
XS Rating Curve= 0 ,0
Exp/Cntr(USF)=0,0
Exp/Cntr=0.3,0.1

Type RM Length L Ch R = 1 ,17221   ,102.4,102.4,102.4
XS GIS Cut Line= 4
2227306.67692772699774.0221537732227478.89106145699763.122525056
2227956.29479924699383.8154457162228250.58477459 699457.93292099
#Sta/Elev= 30
       0 1915.33    53.6 1895.08   121.7 1872.93   141.9 1863.97   161.8 1850.67
     210 1847.79  243.53 1829.59   248.9 1825.09   254.6 1824.04   312.1 1824.14
   331.4 1833.05   345.7 1829.89   368.3  1832.8   394.1 1830.14   409.2 1824.23
   475.6 1824.63  488.721830.126   511.4  1840.9   613.3 1841.41   639.1  1837.2
   659.5 1837.44   720.8 1848.01   786.3 1849.19   811.1 1847.48     836 1855.38
   888.8 1862.46   964.6 1876.82   987.6 1883.36  1000.8 1884.34  1085.8 1914.16
#Mann= 5 ,-1,0
       0      .1       0  243.53    .045       0  488.72     .08       0
  592.56     .06       0   932.3      .1       0
Bank Sta=243.53,488.72
XS Rating Curve= 0 ,0
Exp/Cntr(USF)=0,0
Exp/Cntr=0.3,0.1

Type RM Length L Ch R = 1 ,17118   ,66.4,66.4,66.4
XS GIS Cut Line= 4
2227278.31418637699939.3871243052227504.28460533699949.550836218
2227811.03536289699535.3327606262228186.00696704699588.094258893
#Sta/Elev= 30
       0 1919.44    41.8 1908.87      90 1893.83     174  1862.7     186 1853.23
   190.1 1851.51   239.5 1850.09   281.4 1845.13   360.8 1842.16   380.8 1834.06
  401.021830.114   420.9 1823.84   555.4 1824.03   574.91830.113   602.4 1837.91
     636  1841.7   723.4 1841.74   783.2 1844.53   819.5 1841.77   839.7 1843.54
   855.9 1848.38   871.8 1848.93   896.3 1853.18   920.5 1858.85   928.6  1863.2
   940.7 1866.56     978 1871.51  1057.9 1894.37  1102.3 1905.61  1120.3 1907.66
#Mann= 4 ,-1,0
       0      .1       0  401.02    .045       0   574.9     .08       0
  841.63      .1       0
Bank Sta=401.02,574.9
XS Rating Curve= 0 ,0
Exp/Cntr(USF)=0,0
Exp/Cntr=0.3,0.1

Type RM Length L Ch R = 1 ,17052   ,191.9,191.9,191.9
XS GIS Cut Line= 4
2227284.10178854699992.748860163 2227545.4130447700005.366266038
2227852.16380226699591.1481904462228179.63682781699636.958677211
#Sta/Elev= 30
       0 1920.92    44.1 1908.64   125.9 1879.62   152.3 1867.89   164.3 1864.15
   180.3 1852.98   228.3  1850.4   261.6 1847.07   386.3 1842.42     401 1840.24
   427.71830.093   435.3 1825.42   446.7 1823.72   568.7 1823.75   575.4 1824.87
  587.341830.092   595.4 1833.61   618.3 1836.24   638.3 1842.04   807.2 1842.39
   828.5  1843.6   861.9  1847.8   892.2 1855.51   914.4 1857.59   946.7 1862.96
   950.7 1864.11   958.8 1869.19  1035.6 1892.04  1088.1 1905.88  1107.7 1912.55
#Mann= 7 ,-1,0
       0      .1       0   427.7    .045       0  587.34     .07       0
  621.62     .08       0  701.62     .07       0  751.62     .08       0
  837.05      .1       0
Bank Sta=427.7,587.34
XS Rating Curve= 0 ,0
Exp/Cntr(USF)=0,0
Exp/Cntr=0.3,0.1

Type RM Length L Ch R = 1 ,16860   ,320.5,320.5,320.5
XS GIS Cut Line= 4
2227197.68064056700061.7723518932227478.89106145700061.772351893
2227965.01450221699917.8972528332228217.88588844699924.437030063
#Sta/Elev= 30
       0 1939.58    30.5  1937.2   122.5 1910.51   178.5 1889.91   234.5 1872.22
   242.5 1868.68   258.5 1857.09   266.5 1853.27   290.9 1852.97   361.8 1845.59
   420.2 1844.34   428.6 1842.85   441.1 1835.55   453.3 1832.31  506.231830.027
   524.1  1823.6   566.6  1823.5   633.6 1823.54   653.51830.027   670.5 1836.45
   728.9 1842.66   753.9 1843.58   803.3    1854   823.4 1864.71   939.4 1902.99
   951.4 1905.31   959.4 1910.99   983.4 1913.36   991.4 1917.92  1041.1 1935.48
#Mann= 5 ,-1,0
       0      .1       0  506.23    .045       0   653.5      .1       0
  731.21     .06       0  828.18      .1       0
Bank Sta=506.23,653.5
XS Rating Curve= 0 ,0
Exp/Cntr(USF)=0,0
Exp/Cntr=0.3,0.1

Type RM Length L Ch R = 1 ,16539   ,472,472,472
XS GIS Cut Line= 3
2227351.60581403700425.3453872822228029.14844976  700236.0876317
2228277.15913943700201.036875489
#Sta/Elev= 30
       0 1902.31    29.7 1890.51    75.3 1877.52   104.4 1865.04   137.6 1862.41
   150.1 1857.34   212.4 1850.12   224.9 1844.24   299.3 1841.89   399.3 1843.94
   415.9 1838.77   432.5 1830.34   446.7 1829.12   457.4 1823.28   569.6  1823.3
  579.361828.887   586.2  1833.7   601.2 1834.81   623.6 1841.11     636 1840.97
   648.5 1846.29   665.1 1849.06     690 1860.83   714.6 1861.27   726.7 1869.37
   761.8 1886.04   815.6 1907.39   831.8 1909.91   917.6 1947.91     954 1966.78
#Mann= 5 ,-1,0
       0      .1       0   446.7    .045       0  579.36      .1       0
     580     .06       0     680      .1       0
Bank Sta=446.7,579.36
XS Rating Curve= 0 ,0
Exp/Cntr(USF)=0,0
Exp/Cntr=0.3,0.1

Type RM Length L Ch R = 1 ,16068   ,553.5,553.5,553.5
XS GIS Cut Line= 3
2227508.85702725 700844.113219762228209.00976429700689.910658518
 2228382.4450543700563.309789389
#Sta/Elev= 30
       0 1887.74    60.7  1869.1      73 1861.05   109.9 1860.14   134.5    1848
   208.2 1841.34   343.4 1841.59   371.1 1838.33   396.6 1831.43   413.11829.702
   421.2 1823.46   425.3 1823.19   515.4 1823.34  527.011829.704   544.1 1833.49
   564.5 1841.48   589.1 1843.75   617.8  1855.9   646.4 1856.96   654.6 1863.37
   669.9 1869.71   679.9 1876.31   703.8 1879.58   716.1 1889.59   725.8 1893.46
   831.4 1914.31   860.6 1922.22   874.3 1923.75   884.3 1928.51   931.7 1945.05
#Mann= 5 ,-1,0
       0      .1       0   413.1    .045       0  527.01      .1       0
     610     .06       0     710      .1       0
Bank Sta=413.1,527.01
XS Rating Curve= 0 ,0
Exp/Cntr(USF)=0,0
Exp/Cntr=0.3,0.1

Type RM Length L Ch R = 1 ,15514   ,456.7,456.7,456.7
XS GIS Cut Line= 2
2227592.77385006701305.3884343172228524.83259019701253.859489415
#Sta/Elev= 30
       0 1905.22    63.5 1880.47    91.5 1867.81    99.6 1865.76   115.6 1853.48
   119.6 1851.94   151.6 1853.88   159.1  1851.6   171.7 1844.38   203.7 1839.88
   275.8 1840.86   283.3 1836.14   291.41827.989   299.9 1823.29   303.9 1822.81
     380 1822.81   393.5 1826.15     408 1827.82     424 1835.56   431.7 1837.47
   468.1 1838.68   516.2 1842.91   536.2 1842.69   552.2 1844.69   584.3 1844.87
   660.7  1851.2   732.5 1859.22   844.7  1869.5   880.7 1876.24   933.5 1881.19
#Mann= 6 ,-1,0
       0      .1       0   291.4    .045       0     408      .1       0
     510     .06       0     610      .1       0     810     .08       0
Bank Sta=291.4,408
XS Rating Curve= 0 ,0
Exp/Cntr(USF)=0,0
Exp/Cntr=0.3,0.1

Type RM Length L Ch R = 1 ,15057   ,412.5,412.5,412.5
XS GIS Cut Line= 2
2227604.23171155701683.7316768332228376.01470915701819.816328096
#Sta/Elev= 30
       0 1901.72     8.1 1899.38    16.2 1895.11    64.9 1862.38    81.2 1856.84
    89.3 1852.67   109.6 1847.26     138 1847.28   146.2 1842.42   158.3 1838.75
     203 1840.11   239.6 1839.15   255.8 1835.83  273.53 1829.17   280.2 1823.62
   284.3 1822.41   365.5 1822.53   369.6 1823.87  377.261829.171   393.9 1832.42
   406.1 1838.83   425.9 1840.01   442.7 1843.11   467.3 1843.61   540.6 1851.19
   609.2 1860.52   657.9 1871.11   694.5 1877.51   747.3 1889.12   783.7 1898.72
#Mann= 6 ,-1,0
       0      .1       0  273.53    .045       0  377.26      .1       0
     410     .06       0     510      .1       0     710     .08       0
Bank Sta=273.53,377.26
XS Rating Curve= 0 ,0
Exp/Cntr(USF)=0,0
Exp/Cntr=0.3,0.1

Type RM Length L Ch R = 1 ,14645   ,658,658,658
XS GIS Cut Line= 3
 2227412.1576653701738.1157932082227516.66285203 701899.16816138
2228141.35523116 702457.57783679
#Sta/Elev= 30
       0 1955.36    28.3 1940.59    48.5 1931.99    94.2 1919.77   151.5  1897.4
   184.8 1888.83   201.6 1882.74     219 1871.46   229.9 1866.02     249 1846.28
   255.4 1843.02     295 1841.95   330.8 1846.03     380 1846.23   411.3 1844.87
   438.1 1842.26   456.61828.917     465 1823.43   470.3 1822.32   541.5 1822.28
   547.2 1822.87  553.431828.912   561.5 1838.19     567 1840.66   666.2  1842.3
   741.2 1846.45   825.2 1857.31   879.2 1867.83   945.3 1876.81  1029.9 1891.84
#Mann= 6 ,-1,0
       0      .1       0   456.6    .045       0  553.43      .1       0
  581.99     .06       0  611.99     .07       0  711.99      .1       0
#XS Ineff= 2 , 0
          329.68 1865.55
Permanent Ineff=
       F       F
Bank Sta=456.6,553.43
XS Rating Curve= 0 ,0
Exp/Cntr(USF)=0,0
Exp/Cntr=0.3,0.1

Type RM Length L Ch R = 1 ,13987   ,629.5,629.5,629.5
XS GIS Cut Line= 2
2227155.57617492701688.4298626272227170.37960025 702626.18073991
#Sta/Elev= 30
       0 1982.11    64.8 1959.84    96.8 1944.55   156.8 1911.04   192.8 1895.68
   208.8 1885.37   228.8 1878.52   280.8  1868.2   308.8 1850.88   340.8 1851.06
   408.8 1842.93   508.8 1839.74   548.8 1836.29   568.8  1830.6   596.8 1832.46
  606.32 1828.49   616.8 1822.12   620.8 1822.06   692.8 1822.06   700.8 1823.79
   707.51828.494   712.8  1832.8   724.8 1838.04   752.8 1842.16   768.8 1852.34
   788.8 1854.19   800.8 1864.71   812.9 1871.54   861.9 1880.49   937.9 1908.23
#Mann= 4 ,-1,0
       0      .1       0  606.32    .045       0   707.5     .07       0
     790      .1       0
Bank Sta=606.32,707.5
XS Rating Curve= 0 ,0
Exp/Cntr(USF)=0,0
Exp/Cntr=0.3,0.1

Type RM Length L Ch R = 1 ,13357   ,614.5,614.5,614.5
XS GIS Cut Line= 4
2226662.08718632701641.3328939142226558.02866582701925.796888775
2226568.99343592702508.4960999992226634.66120765702726.644471852
#Sta/Elev= 30
       0  1925.5     123 1889.49   170.2 1879.32   234.1 1869.23   263.9 1860.42
   276.7 1860.99   293.7 1854.18   314.3 1849.42   326.3 1843.72   362.3 1845.13
   422.2 1840.09   506.3 1842.59   523.71827.938   530.3 1824.59   546.3 1821.88
   610.3 1821.88   614.3 1822.55  622.131827.892   646.3 1828.63   674.3 1835.19
   774.4 1840.13   814.4 1844.27   846.4 1848.91   878.4 1858.22   903.1 1859.05
   928.2 1868.92   974.1  1874.6     995 1885.43  1024.3 1890.85  1113.5  1918.5
#Mann= 7 ,-1,0
       0      .1       0   523.7    .045       0  622.13      .1       0
   662.9     .07       0   752.9     .05       0   852.9     .07       0
   955.7      .1       0
Bank Sta=523.7,622.13
XS Rating Curve= 0 ,0
Exp/Cntr(USF)=0,0
Exp/Cntr=0.3,0.1

Type RM Length L Ch R = 1 ,12743   ,597.3,597.3,597.3
XS GIS Cut Line= 2
2225745.12284916702143.8235649952226365.25394419702836.113867624
#Sta/Elev= 30
       0 1975.05    16.6 1970.52    59.8 1950.84    79.6  1940.3   113.6 1926.49
   190.1  1892.3   205.9 1882.84   216.6 1880.75   232.7 1872.79     265 1859.88
   286.4 1846.48     326  1844.2   334.3 1841.72  349.541827.363   354.4 1823.63
   361.6 1821.72     445 1821.88   457.81827.364   490.5 1834.92   565.7 1839.35
   640.9 1841.95   654.6 1844.77   673.1 1845.77     730 1856.36     768 1857.45
   789.9 1866.38   841.6  1870.2   861.9 1874.72   898.6 1890.74   929.4 1902.37
#Mann= 6 ,-1,0
       0      .1       0  349.54    .045       0   457.8      .1       0
     730     .06       0     840     .07       0     880      .1       0
Bank Sta=349.54,457.8
XS Rating Curve= 0 ,0
Exp/Cntr(USF)=0,0
Exp/Cntr=0.3,0.1

Type RM Length L Ch R = 1 ,12146   ,497.8,497.8,497.8
XS GIS Cut Line= 4
2225392.17218533702581.460914694 2225442.7549067 702713.69394051
2225860.98256637703142.8863702822226126.82863319703175.104434687
#Sta/Elev= 30
       0 1929.14   119.6 1878.58   146.4 1855.76   185.5 1856.52   213.5 1842.28
   281.2 1834.37  301.271826.871   308.4 1822.18     314 1821.41   402.5 1821.42
  420.211826.874   430.2 1828.45   447.7 1837.32   464.7 1842.84     558 1838.17
   569.3 1840.18     592 1839.56   665.2 1845.36   722.5 1847.55   740.8 1852.11
   764.2 1854.76   840.8 1855.65   848.8 1859.02   882.3 1863.07   905.2 1863.86
   914.7 1868.81   932.6 1874.68   957.6 1877.56   973.7 1886.24  1008.6 1893.38
#Mann= 4 ,-1,0
       0      .1       0  301.27    .045       0  420.21      .1       0
  820.84     .06       0
Bank Sta=301.27,420.21
XS Rating Curve= 0 ,0
Exp/Cntr(USF)=0,0
Exp/Cntr=0.3,0.1

Type RM Length L Ch R = 1 ,11648   ,611.3,611.3,611.3
XS GIS Cut Line= 3
2224913.87561894703366.9833568652225054.28876589703263.498841422
 2226136.5289732703215.940984476
#Sta/Elev= 30
       0 1887.52      83 1865.96   168.9 1849.06   236.4  1842.6   280.4 1840.66
   332.5  1841.2   340.5 1835.08  346.361826.368     351  1822.1   356.5 1821.31
   444.6 1821.31   448.6 1822.56  451.771826.364   456.6 1828.69   484.6 1830.07
   508.6 1837.01   520.6 1838.65   636.8 1840.12   684.7 1838.53   752.9 1839.23
     893  1845.4     909 1848.59   953.1 1848.91   965.1  1851.9   985.1  1852.1
  1073.2 1863.09  1125.2 1865.03  1137.2 1870.34  1173.3 1873.41  1257.7  1891.6
#Mann= 5 ,-1,0
       0      .1       0  346.36    .045       0  451.77      .1       0
 1064.43     .06       0 1254.43      .1       0
Bank Sta=346.36,451.77
XS Rating Curve= 0 ,0
Exp/Cntr(USF)=0,0
Exp/Cntr=0.3,0.1

Type RM Length L Ch R = 1 ,11036   ,541.5,541.5,541.5
XS GIS Cut Line= 2
2225311.91851826703900.8960196662226059.91482397703396.642478396
#Sta/Elev= 30
       0 1877.05    34.1  1871.1    60.5    1863    80.7 1861.94   125.7 1852.17
   188.4  1842.7   260.8 1838.22   365.9 1837.17   405.5 1834.27   449.7 1825.86
   458.1 1821.49   463.4 1820.76   521.3 1820.72     572 1820.72   584.71825.859
   590.7 1827.94   603.3 1836.84   636.4 1840.34     657 1844.38   675.7  1845.5
   697.3 1850.32   717.5  1850.9   746.3  1859.9   767.3 1872.67   775.1 1875.53
   812.6 1880.69   839.7 1882.22   854.2 1885.61   873.5 1885.51   902.1 1889.48
#Mann= 7 ,-1,0
       0      .1       0   449.7    .045       0   584.7      .1       0
     640     .06       0     760      .1       0     800     .06       0
     870      .1       0
Bank Sta=449.7,584.7
XS Rating Curve= 0 ,0
Exp/Cntr(USF)=0,0
Exp/Cntr=0.3,0.1

Type RM Length L Ch R = 1 ,10495   ,564.3,564.3,564.3
XS GIS Cut Line= 2
2225629.79043582704255.3630018912226391.72803082703881.841884419
#Sta/Elev= 30
       0 1876.18    69.2 1860.09   109.6 1852.82   204.9 1840.68   229.8 1840.28
   293.4  1830.7   323.4 1834.35   341.2 1828.13  344.281825.483   350.1 1820.66
   358.7 1820.25   461.5 1820.25     466 1820.59  471.231825.485   477.5 1831.44
   483.8 1833.37   528.3 1835.07   537.2 1837.93   556.4 1837.89   583.3 1841.52
   595.6  1844.7   626.3 1847.26   648.6 1851.82     662  1857.6   675.3  1859.8
     711 1870.39   729.8 1878.27   742.2 1879.98   750.7 1884.91   848.6 1923.73
#Mann= 4 ,-1,0
       0      .1       0  344.28    .045       0  471.23     .06       0
     560      .1       0
Bank Sta=344.28,471.23
XS Rating Curve= 0 ,0
Exp/Cntr(USF)=0,0
Exp/Cntr=0.3,0.1

Type RM Length L Ch R = 1 ,9931    ,652.2,652.2,652.2
XS GIS Cut Line= 2
2226207.56408941 704756.988985532226546.43390963704153.326991251
#Sta/Elev= 30
       0 1893.79    13.5 1887.75    22.7 1887.73    29.7 1886.13    44.4 1879.08
    59.1 1873.47     119 1853.67   176.6 1838.51   183.3 1835.95   206.2 1834.33
   211.8 1831.75  217.981824.989   220.7 1821.79   223.6 1820.17   229.1 1819.91
   320.5 1819.92  334.021824.983   352.9 1827.59   366.8 1831.39   388.1 1831.37
     394 1833.35   409.8  1836.3   490.9  1838.8   508.6 1840.58   532.4 1845.94
   568.6 1849.01   600.7 1858.41   609.9  1862.2   628.2 1866.34   692.3 1892.15
#Mann= 4 ,-1,0
       0      .1       0  217.98    .045       0  334.02     .06       0
     480      .1       0
Bank Sta=217.98,334.02
XS Rating Curve= 0 ,0
Exp/Cntr(USF)=0,0
Exp/Cntr=0.3,0.1

Type RM Length L Ch R = 1 ,9278    ,559.6,559.6,559.6
XS GIS Cut Line= 2
2226820.32660308705027.7586374592227121.26436116704333.739631578
#Sta/Elev= 30
       0 1914.26    50.8  1891.7    68.2 1879.84    80.9 1878.97      84 1877.68
   103.1 1865.89   124.9 1854.38   172.8  1830.9   199.5 1829.79   212.1 1826.74
  215.641824.618   225.2 1819.55   238.2 1818.31   329.8 1818.49  344.53 1824.62
   360.3 1832.05   364.7 1833.04   390.8 1833.09   418.5 1831.24   447.5  1836.3
   500.6 1836.94   543.4 1841.84   560.9 1842.57   588.8 1848.29   600.1 1851.99
     613 1852.16     635 1861.18   670.9 1871.03   698.3 1880.22   756.5 1902.42
#Mann= 4 ,-1,0
       0      .1       0  215.64    .045       0  344.53     .06       0
     430      .1       0
Bank Sta=215.64,344.53
XS Rating Curve= 0 ,0
Exp/Cntr(USF)=0,0
Exp/Cntr=0.3,0.1

Type RM Length L Ch R = 1 ,8719    ,654.6,654.6,654.6
XS GIS Cut Line= 2
2227233.02621835705301.2759634042227727.98141747704588.380390338
#Sta/Elev= 30
       0  1932.4    48.3 1910.36    87.8 1893.44    96.7 1890.95   110.7 1883.32
   121.9  1874.8   140.3 1872.23     169 1855.57   194.9 1844.06   212.1 1838.72
   224.1 1836.88   229.4 1833.99   263.9 1834.57   286.9 1832.19   307.1 1827.22
   321.5 1825.99  323.891824.414   331.2 1819.15     341 1817.47   433.4 1817.47
  441.91 1824.41   457.9 1834.01   462.2 1835.15   491.9 1835.96   671.8 1847.78
   764.6 1857.71   812.1 1867.11   833.1 1868.07   861.2  1872.4   867.9 1874.75
#Mann= 6 ,-1,0
       0      .1       0  323.89    .045       0  441.91      .1       0
     450     .06       0     570     .05       0     660      .1       0
Bank Sta=323.89,441.91
XS Rating Curve= 0 ,0
Exp/Cntr(USF)=0,0
Exp/Cntr=0.3,0.1

Type RM Length L Ch R = 1 ,8064    ,738.2,738.2,738.2
XS GIS Cut Line= 3
2227504.31625065705643.9973596212227769.17528331705582.771252475
 2228223.1167656705147.156600214
#Sta/Elev= 30
       0 1915.91    62.3 1893.48    88.9 1873.53    98.4 1869.48   135.3 1869.09
   147.7 1872.37   205.1  1856.4   246.2 1848.56   306.2 1839.93   348.6 1835.94
   422.2 1835.38   435.9 1830.16   447.7 1822.71   473.1 1823.55   482.1 1818.29
   487.9 1817.03     563 1817.22   574.6 1819.13  583.791823.484   603.3 1831.21
   620.8 1834.57   682.5 1835.17   702.9 1839.18   725.1 1839.37   736.1 1845.05
   782.5 1855.33   795.6 1861.31   818.3 1862.62   851.9 1876.34     901 1892.33
#Mann= 5 ,-1,0
       0      .1       0   473.1    .045       0  583.79      .1       0
  641.84     .06       0  731.84      .1       0
Bank Sta=473.1,583.79
XS Rating Curve= 0 ,0
Exp/Cntr(USF)=0,0
Exp/Cntr=0.3,0.1

Type RM Length L Ch R = 1 ,7326    ,576,576,576
XS GIS Cut Line= 2
2227529.51673675705987.3712693012228388.05823587706125.527372607
#Sta/Elev= 30
       0 1894.47    35.1 1883.71    51.3 1876.04    63.5 1874.08     108 1859.48
   128.3 1856.24   148.5 1862.27   164.8 1861.75   189.3 1845.87   205.3  1840.3
   302.5 1834.98   432.1 1833.89   472.7 1836.97   506.4 1825.77   529.4 1825.85
  533.52 1823.86   545.6 1816.75   638.8 1816.75   642.8 1818.23  646.351823.859
   663.1 1834.98   679.3 1836.11   683.3 1838.38   703.6 1861.79   727.9 1868.26
   754.2 1893.88   784.6 1910.33   796.8 1913.21   825.1 1930.51   869.6 1948.75
#Mann= 5 ,-1,0
       0      .1       0  533.52    .045       0  646.35     .05       0
     680     .06       0     780      .1       0
Bank Sta=533.52,646.35
XS Rating Curve= 0 ,0
Exp/Cntr(USF)=0,0
Exp/Cntr=0.3,0.1

Type RM Length L Ch R = 1 ,6750    ,228.6,228.6,228.6
XS GIS Cut Line= 4
2227470.47758148706133.4017709252227709.96552475706225.620059696
2227786.09235718706621.7615395842227995.40923181706703.668058182
#Sta/Elev= 30
       0 1892.14      79 1868.77    91.8 1862.73   186.1 1844.86   224.7  1842.9
   256.6 1858.24   406.9 1857.74     415  1854.1   419.1 1838.12   423.2 1826.94
  457.981823.684     468 1817.45   480.2  1816.5   565.7  1816.5   579.11823.682
   586.1 1826.82   602.4 1827.53   606.5  1833.5   610.5 1848.65   614.6 1857.78
   618.7 1858.91   651.1  1858.7   666.6 1853.38     688 1842.55     761 1839.53
   786.8    1843   816.9 1859.52   849.5 1864.43   861.8 1872.63   884.8 1881.78
#Mann= 4 ,-1,0
       0      .1       0  457.98    .045       0   579.1     .06       0
  680.02      .1       0
Bank Sta=457.98,579.1
XS Rating Curve= 0 ,0
Exp/Cntr(USF)=0,0
Exp/Cntr=0.3,0.1

Type RM Length L Ch R = 1 ,6521    ,168.7,168.7,168.7
XS GIS Cut Line= 3
2227389.78135139706509.3030759152227788.97773471706755.631125634
2227940.47761793706796.198425492
#Sta/Elev= 30
       0 1880.73     7.5 1879.38    45.1 1866.24   120.3 1845.09   167.3 1836.53
   190.8 1835.19   196.4 1832.64  204.511823.574   209.6 1820.26   223.7 1816.31
   298.9  1816.5  312.511823.577   322.4 1824.62   342.5 1824.16   369.4 1831.74
   402.3 1833.26   430.5 1840.74     454 1840.47   493.1 1855.57   505.5 1858.87
   530.4 1859.53   541.5 1855.99   551.1 1855.17   555.2 1855.71   563.5  1859.8
   567.5 1860.39   604.9 1861.58     609 1862.88   621.5 1873.01   625.9 1875.14
#Mann= 5 ,-1,0
       0      .1       0  204.51    .045       0  312.51     .07       0
     380     .06       0  489.08      .1       0
Bank Sta=204.51,312.51
XS Rating Curve= 0 ,0
Exp/Cntr(USF)=0,0
Exp/Cntr=0.3,0.1

Type RM Length L Ch R = 1 ,6353    ,24,24,24
XS GIS Cut Line= 3
2227295.38655467706771.7903940632227372.20208916706812.697990411
2227921.46260217706814.702826004
#Sta/Elev= 30
       0 1874.18    23.6 1867.62    32.6 1862.93    75.5 1848.39     103  1841.9
     139 1835.72     171 1834.39     235 1835.56     239 1832.22  242.981823.514
     247 1819.93     251 1818.68     259 1816.59   266.8 1816.19     331 1816.19
     335 1816.56     347 1822.63  376.861823.506     383  1826.5     387 1833.35
     391 1835.34     487 1836.49     503 1842.89     511  1847.5   524.1 1857.28
     531 1859.88     567 1859.02   596.4 1859.95     631 1861.87   636.3 1864.78
#Mann= 6 ,-1,0
       0      .1       0  242.98    .045       0  376.86     .07       0
  427.03     .06       0  527.03     .07       0  627.03      .1       0
Bank Sta=242.98,376.86
XS Rating Curve= 0 ,0
Exp/Cntr(USF)=0,0
Exp/Cntr=0.3,0.1

Type RM Length L Ch R = 1 ,6329    ,217.6,217.6,217.6
XS GIS Cut Line= 3
2227286.61357989706810.1945136992227357.36788517706836.972142384
2227918.08388338706837.598459657
#Sta/Elev= 30
       0 1870.15    31.6 1860.29    61.5 1848.82    94.5 1840.08   126.5 1834.74
   138.5 1833.92   218.5 1834.38   222.5 1833.82   234.5 1829.03  243.471823.507
   246.5 1820.24   250.4 1818.75   270.4 1816.16   338.5 1816.16   354.5 1821.99
   370.5 1822.06  379.091823.507   382.5 1824.25   386.5 1826.85   390.5 1831.66
   398.6 1834.52   474.2  1836.4   494.5 1834.99   510.5 1842.33   518.5  1847.1
   530.8 1856.38   538.8 1859.85   626.5 1861.57   630.5 1862.51   636.4 1865.87
#Mann= 6 ,-1,0
       0      .1       0  243.47    .045       0  379.09     .07       0
  425.65     .06       0  525.65     .07       0  625.65      .1       0
Bank Sta=243.47,379.09
XS Rating Curve= 0 ,0
Exp/Cntr(USF)=0,0
Exp/Cntr=0.3,0.1

Type RM Length L Ch R = 1 ,6111    ,444.6,444.6,444.6
XS GIS Cut Line= 3
2227228.16026491706899.3842911312227755.14358696707167.279923241
2227999.97998929707136.927569177
#Sta/Elev= 30
       0 1875.69      18 1868.65    26.9 1867.04    80.8 1845.48   107.7 1838.91
   134.6 1833.54     175 1834.47     193 1832.88   206.4 1825.05   218.5 1823.12
   230.4 1823.39   239.3  1817.1   246.8 1815.69   332.1 1815.69   340.5  1817.8
  350.251823.448   363.5 1831.51   383.5 1836.46   453.5  1835.6   551.9 1838.72
   616.4 1846.83   652.7 1855.88   672.8 1856.19   680.9 1861.27     697 1866.54
   713.1 1860.19   741.3 1861.15   753.4 1867.63   777.6 1886.08   837.9 1905.25
#Mann= 5 ,-1,0
       0      .1       0   230.4    .045       0  350.25      .1       0
     540     .06       0  641.17      .1       0
Bank Sta=230.4,350.25
XS Rating Curve= 0 ,0
Exp/Cntr(USF)=0,0
Exp/Cntr=0.3,0.1

Type RM Length L Ch R = 1 ,5667    ,837.9,837.9,837.9
XS GIS Cut Line= 4
2226809.26130083707013.1341176062227047.81326075707403.107989768
 2227794.6193489 707488.983295122228017.68483886707349.694063129
#Sta/Elev= 30
       0 2002.66    36.2 1982.53    77.8    1964   112.6 1956.28   165.1 1938.71
   310.5 1897.64   481.7 1858.02   517.9 1841.84   542.1 1833.78   618.6 1830.53
   647.1  1822.6   658.8 1815.92   662.9 1815.66   767.5 1815.66   771.6 1816.68
   777.1 1822.75   787.7 1828.79   827.7 1836.32   884.3 1834.11  1021.2 1834.36
  1154.1 1838.13  1267.3 1846.53  1300.3  1853.3  1323.1 1853.44  1356.9 1863.89
  1369.5 1859.82  1395.7 1859.47  1421.8 1873.43  1442.1 1877.11  1471.9  1886.7
#Mann= 5 ,-1,0
       0      .1       0   647.1    .045       0   777.1      .1       0
 1338.88     .06       0 1458.88      .1       0
Bank Sta=647.1,777.1
XS Rating Curve= 0 ,0
Exp/Cntr(USF)=0,0
Exp/Cntr=0.3,0.1

Type RM Length L Ch R = 1 ,4829    ,596.9,596.9,596.9
XS GIS Cut Line= 3
2227532.43174357708606.7701440612227826.66257997707526.381485332
2228104.21190632707395.273850386
#Sta/Elev= 30
       0 2070.11    30.7  2071.3    51.4 2066.06   101.1 2037.27   159.2  1997.8
   213.4 1965.16   320.9 1921.03   395.3 1882.99   519.9 1838.54   540.6    1834
   569.6 1832.75   577.9 1829.61   583.71823.484   594.5 1815.08   606.9 1814.94
     694 1815.01   718.71822.991   734.2  1823.4   763.5 1831.02   843.2 1829.15
  1122.6 1842.92  1178.9 1848.15    1201 1853.26  1218.7 1852.81  1249.7 1863.25
  1258.5 1859.54  1289.5 1859.58  1298.4 1863.52  1311.6 1873.39  1426.7 1902.25
#Mann= 6 ,-1,0
       0      .1       0   583.7    .045       0   718.7    .025       0
     750      .1       0 1209.74     .06       0 1319.74      .1       0
Bank Sta=583.7,718.7
XS Rating Curve= 0 ,0
Exp/Cntr(USF)=0,0
Exp/Cntr=0.3,0.1

Type RM Length L Ch R = 1 ,4232    ,685.4,685.4,685.4
XS GIS Cut Line= 4
2228020.48656663708553.9740648562228161.21376655708443.013060136
2228346.86066778707965.3590538562228483.99825229707816.201835387
#Sta/Elev= 30
       0 1907.97    65.9 1879.69   101.5 1867.68   126.9  1856.6     137  1855.6
   172.8 1842.86   198.4 1836.84   301.3 1828.93   331.4 1823.88   364.1 1823.12
   395.8 1828.37   411.6 1823.22   463.4 1814.47   571.7 1814.47     576 1815.94
  583.391823.156   640.5 1830.23     665 1830.97   687.6 1842.61   709.7 1857.18
     738 1857.66   740.9 1858.57   752.7 1869.02   784.3 1878.77     800 1885.83
   831.4 1889.34   854.1 1887.95   859.8    1890   870.9 1897.88   894.3 1904.33
#Mann= 4 ,-1,0
       0      .1       0   411.6    .045       0  583.39     .06       0
  679.21      .1       0
Bank Sta=411.6,583.39
XS Rating Curve= 0 ,0
Exp/Cntr(USF)=0,0
Exp/Cntr=0.3,0.1

Type RM Length L Ch R = 1 ,3546    ,734.3,734.3,734.3
XS GIS Cut Line= 3
 2228536.7378181708958.1712969782229039.24788312708234.481718454
2229076.43007041708006.184829004
#Sta/Elev= 30
       0 1888.01      45 1870.99    93.7 1855.96   141.1 1843.28     196 1833.45
   273.9 1824.94   350.9 1830.05   426.8  1829.5   454.4 1826.37   478.4 1819.69
   502.61820.996   514.8  1815.2   520.5 1814.44   630.2 1814.44   634.3 1816.18
   637.51820.685   648.9 1831.97   652.7 1833.63     716 1834.57   830.9  1857.9
   843.7 1856.61   876.9 1858.37   886.5 1862.65   898.6 1871.87   955.3 1888.18
   983.7 1888.71   995.8 1895.42  1044.5 1909.69  1056.6 1911.16  1112.4  1934.4
#Mann= 6 ,-1,0
       0      .1       0   502.6    .045       0   637.5     .06       0
     710      .1       0     790     .06       0     830      .1       0
Bank Sta=502.6,637.5
XS Rating Curve= 0 ,0
Exp/Cntr(USF)=0,0
Exp/Cntr=0.3,0.1

Type RM Length L Ch R = 1 ,2812    ,552.7,552.7,552.7
XS GIS Cut Line= 2
2229033.43444173709251.6232492852229800.19010032708629.887207014
#Sta/Elev= 30
       0 1874.48    39.6 1857.87    54.7  1854.6   103.2 1836.22   127.1 1829.88
   145.9  1828.1     1531822.991   160.1 1815.28   168.3 1813.75   270.6 1813.75
   276.7 1815.33   284.21822.991   290.9 1826.02   307.4 1828.28   358.9 1831.98
   420.7 1832.16   509.9 1829.73   586.7  1830.8     635 1829.82   647.2 1830.94
   678.1 1837.48   755.4 1841.42     776 1841.08   782.9 1843.12   797.7 1853.62
   848.3 1861.48   894.4 1862.79   913.7 1871.09   936.5 1873.86   987.2 1884.57
#Mann= 6 ,-1,0
       0      .1       0     153    .045       0   284.2      .1       0
     450     .05       0     610     .06       0     700      .1       0
Bank Sta=153,284.2
XS Rating Curve= 0 ,0
Exp/Cntr(USF)=0,0
Exp/Cntr=0.3,0.1

Type RM Length L Ch R = 1 ,2259    ,341.8,341.8,341.8
XS GIS Cut Line= 2
2229363.21995019709616.8028852072230001.47138203709291.410967066
#Sta/Elev= 30
       0  1883.4    43.2 1861.47    54.9 1852.43    65.9 1849.88    86.7 1838.61
    99.8 1833.64   158.2 1827.95   176.2 1823.32   196.7 1820.78   211.6 1813.87
   216.6 1813.62   315.4 1813.62   319.9  1814.9  323.871820.927   333.3 1826.61
   339.4 1827.85   351.3 1826.38   369.2 1817.99   378.1 1817.22   413.8 1827.14
   508.4  1831.2   539.9  1834.8   565.4 1840.24   589.3 1841.07   616.2 1850.14
   634.1 1850.16   670.1    1858     688 1862.73   705.2 1871.24   716.4 1871.94
#Mann= 6 ,-1,0
       0      .1       0   196.7    .045       0  323.87      .1       0
     350     .06       0     460     .07       0     580      .1       0
Bank Sta=196.7,323.87
XS Rating Curve= 0 ,0
Exp/Cntr(USF)=0,0
Exp/Cntr=0.3,0.1

Type RM Length L Ch R = 1 ,1917    ,286.1,286.1,286.1
XS GIS Cut Line= 2
2229432.07992111  709831.65055682230135.07958869709815.060594143
#Sta/Elev= 30
       0 1867.32    16.1 1861.32    36.1 1859.64    80.1 1839.11   100.1  1831.3
   148.1 1828.81   172.1 1824.03   178.4 1820.02   188.1 1814.26   196.1 1813.53
   300.2 1813.53   304.2 1814.31  310.49 1820.05   320.2 1826.66   328.2 1827.89
   344.2 1824.85   360.2 1823.97   432.5 1826.21   452.2 1828.16   464.2 1831.93
   500.2 1837.74   516.2 1842.96   544.2 1845.06   564.3 1852.19   584.3 1854.96
   632.3  1866.5   664.3 1880.59   692.3 1882.02   696.3 1883.45   703.2 1889.34
#Mann= 5 ,-1,0
       0      .1       0   178.4    .045       0  310.49      .1       0
     440     .06       0     540      .1       0
Bank Sta=178.4,310.49
XS Rating Curve= 0 ,0
Exp/Cntr(USF)=0,0
Exp/Cntr=0.3,0.1
