--- MIDFKRV2.prj (project) ---

Proj Title=MIDFKRV2
Current Plan=p01
Default Exp/Contr=0,0
English Units
Geom File=g01
Flow File=f01
Plan File=p01
BEGIN DESCRIPTION:
END DESCRIPTION:
DSS Export Rating Curves= 0
DSS Export Rating Curve Sorted= 0
DSS Export Volume Flow Curves= 0
DXF OffsetX= 0
DXF OffsetY= 0
DXF ScaleX= 0
DXF ScaleY= 0

--- MIDFKRV2.p01 (plan) ---

Plan Title=Floodplain
Program Version=4.00
Geom File=g01
Flow File=f01
K Sum by GR=0
Std Step Tol=0.01
Critical Tol=0.01
Num of Std Step Trials=20
Max Error Tol=0.3
Flow Tol Ratio=0.001
Split Flow NTrial=30
Split Flow Tol=0.02
Split Flow Ratio=0.02
Log Output Level=0
Friction Slope Method=1
Unsteady Friction Slope Method=2
Unsteady Bridges Friction Slope Method=1
Global Log Level=0
CheckData=False
Run HTab=0
Run UNet=0
Run PostProcess=0
UNET Theta=0
UNET Theta Warmup=0
UNET ZTol=0
UNET ZSATol=0
UNET MxIter=0
UNET MaxInSteps=0
UNET DtIC=0
UNET DtMin=0
UNET MaxCRTS=0
UNET WFStab=0
UNET SFStab=0
UNET WFX=0
UNET SFX=0
UNET DSS MLevel=0
UNET DZMax Abort=0
UNET Convert EG Bridges=0
UNET Use Existing IB Tables=0
UNET Froude Limit=0
UNET Froude Power=0
Write IC File=0
Echo Input=False
Echo Output=False
Write Detailed=0

--- MIDFKRV2.f01 (steady flow) ---

Flow Title=NFF Regression Equation
Program Version=4.10
Number of Profiles= 1
Profile Names=P100yr
River Rch & RM=MIDFKRV2,Main            ,73015.9
15704.47
River Rch & RM=MIDFKRV2,Main            ,214.3
   17181
River Rch & RM=MIDFKRV2,Main            ,214.3
17179.22
Boundary for River Rch & Prof#=MIDFKRV2,Main            , 1
Up Type= 0
Dn Type= 3
Dn Slope=0.025
DSS Import GetInterval= 0
DSS Import GetPeak= 0
DSS Import FillOption= 0

--- MIDFKRV2.g01 (geometry) ---

Geom Title=USGS 10m DEM
Program Version=4.10

River Reach=MIDFKRV2        ,Main
Reach XY= 30
     1802521.636      163237.718     1801996.071      163729.777
     1802940.711      164783.142     1805336.544       164744.08
      1805894.27      165974.548     1808205.468      167445.903
     1808123.002      168717.604     1805657.182      169491.982
     1805724.022      171122.624     1807115.949      170539.291
     1808808.658      173549.708     1811402.895      173613.001
     1811705.793      180440.333      1813071.45      181345.691
     1810822.981      183303.614     1810812.495      184538.564
     1813805.644      186691.853     1811300.629      188212.363
     1809679.752      190587.468     1811156.314      192774.968
     1810724.022       196082.26     1808977.691      195053.429
     1807038.632      197278.969     1808735.741      197962.468
     1808087.304      200097.885     1809720.116      200784.083
     1811668.033      200312.728     1812401.106      201039.291
     1811317.772      204237.208     1813149.044      205061.396

Type RM Length L Ch R = 1 ,73015.9 ,1279.8,1228.1,1176.3
XS GIS Cut Line= 3
      1802106.46      162691.842     1802783.543      163655.384
     1802942.758       163755.63
#Sta/Elev= 30
       0 2086.83    78.5 2066.39    98.1 2060.16   147.2 2041.22   235.5 2003.22
   304.2 1978.28   323.8  1969.9   372.9 1945.05   392.6 1938.13     422 1930.32
   431.8 1926.55   451.4 1916.84   490.7 1893.33   539.8    1867   608.4 1826.55
   618.3 1822.36   628.1 1820.84   637.9 1820.79   706.6  1820.8   716.4 1821.26
   726.2 1823.22   755.7 1833.16   765.5  1834.4  785.541834.788   902.9 1836.97
 1111.251837.111  1128.6 1839.12 1153.761844.332  1318.8 1878.24  1365.8 1888.71
#Mann= 6 ,-1 , 0
       0     .12       0   618.3    .045       0   726.2    .016       0
  785.54     .12       0 1111.25     .06       0 1153.76     .12       0
#XS Ineff= 2 , 0
                          940.98          1930.5
Permanent Ineff=
       F       F
Bank Sta=618.3,726.2
XS Rating Curve= 0 ,0
Exp/Cntr=0.3,0.1

Type RM Length L Ch R = 1 ,71787.8 ,474.1,468.4,463.1
XS GIS Cut Line= 3
     1801630.015      164370.326     1802672.583      163896.878
     1802867.441      163878.021
#Sta/Elev= 30
       0 2084.33    39.2 2081.44    58.7 2078.32    97.9  2063.2     137 2045.75
   225.1 2001.44   244.7  1992.4   283.8 1975.53   352.3 1950.42   420.8 1914.63
   479.5 1889.94  533.221868.862  573.461853.908   606.8 1841.04   616.6 1838.99
   645.9 1838.14   665.5  1834.9   675.3 1831.73  699.211821.497   704.6 1819.82
   724.2 1818.95   792.7  1821.5  831.841824.632   861.2 1829.18  891.82 1829.39
  896.24 1829.39   998.2 1831.49  1096.1 1841.79  1174.4 1852.72  1340.8 1881.43
#Mann= 8 ,-1 , 0
       0     .12       0  533.22    .016       0  573.46     .12       0
  699.21    .045       0   792.7     .12       0  831.84    .016       0
  891.82     .06       0  896.24     .12       0
Bank Sta=699.21,792.7
XS Rating Curve= 0 ,0
Exp/Cntr=0.3,0.1

Type RM Length L Ch R = 1 ,71319.4 ,450.5,442.4,432.2
XS GIS Cut Line= 3
     1802072.733      164759.582     1802606.795      164390.135
      1802916.04      164207.976
#Sta/Elev= 30
       0 1971.18    88.6 1943.44   216.5 1902.64   295.2 1873.91   314.9 1868.14
  368.371854.503  396.511846.597   432.9 1838.91   462.4 1833.73   482.1 1833.01
   619.9 1832.09   629.7 1830.69   639.6 1826.79   649.4 1820.89  654.961818.855
   659.1 1817.34   668.8 1816.73   688.2 1817.02   746.4 1819.66   756.1 1821.47
   765.8  1825.7   775.5 1830.98  777.661831.753   785.2 1834.45  809.151838.218
   843.4 1844.49  880.431849.583   901.6 1852.85  928.621858.407  1008.3 1877.51
#Mann= 9 ,-1 , 0
       0     .12       0  368.37    .016       0  396.51     .12       0
  654.96    .045       0   746.4     .12       0  777.66    .016       0
  809.15     .12       0  880.43    .016       0  928.62     .12       0
Bank Sta=654.96,746.4
XS Rating Curve= 0 ,0
Exp/Cntr=0.3,0.1

Type RM Length L Ch R = 1 ,70877.1 ,505.6,482.7,461.6
XS GIS Cut Line= 3
     1802565.531      165040.461     1802895.889      164728.122
      1803162.19      164447.765
#Sta/Elev= 30
       0 1905.56    77.4  1890.6   164.4 1870.54   212.8 1860.51  241.951852.885
  279.421841.196   290.2 1838.09   299.9 1835.89   309.5 1834.47   367.6 1828.86
   377.2 1827.13   386.9 1824.36   406.3 1817.96   415.9 1816.83   425.6 1816.68
   464.3 1816.88  504.421818.732   512.6 1819.55   522.3  1821.8  531.151825.614
   541.6  1829.8   551.3 1831.98  573.071834.008   628.6  1839.9   667.3 1841.05
   696.3 1844.64   725.3 1849.57   754.3 1855.36     822  1869.5   841.3 1874.71
#Mann= 7 ,-1 , 0
       0     .12       0  241.95    .016       0  279.42     .12       0
   406.3    .045       0  504.42     .12       0  531.15    .016       0
  573.07     .12       0
Bank Sta=406.3,504.42
XS Rating Curve= 0 ,0
Exp/Cntr=0.3,0.1

Type RM Length L Ch R = 1 ,70394.3 ,474.3,465.9,457.5
XS GIS Cut Line= 2
     1803242.978      165265.314     1803396.981      164532.126
#Sta/Elev= 30
       0 1922.01    29.2 1908.25    77.8  1886.9     107 1875.18     1481859.968
   165.4 1853.94   184.9 1847.64  198.46 1842.63     253  1821.1   262.7 1818.05
   272.4 1816.88   291.9 1816.68   340.5 1816.69   350.3 1816.82  354.051817.199
     360  1817.8   369.7 1820.12  386.691824.803   398.9    1827  418.341828.147
   496.2 1834.37   583.8 1840.71   622.7 1843.01   632.4 1844.05   642.2 1845.61
   651.9 1847.63   671.4 1852.27   690.8 1857.54   729.7 1869.38   749.2  1874.7
#Mann= 7 ,-1 , 0
       0     .12       0     148    .016       0  198.46     .12       0
   272.4    .045       0  354.05     .12       0  386.69    .016       0
  418.34     .12       0
Bank Sta=272.4,354.05
XS Rating Curve= 0 ,0
Exp/Cntr=0.3,0.1

Type RM Length L Ch R = 1 ,69928.5 ,426.1,424.7,423.4
XS GIS Cut Line= 3
     1803778.979      165336.571     1803772.151      164909.801
     1803762.589      164494.904
#Sta/Elev= 30
       0 1930.15    48.5 1909.11   116.4 1882.51   145.5  1871.8  210.651849.173
   244.21838.571   271.6 1831.94   300.7 1826.01   320.1 1820.54   329.8 1818.46
   339.5 1817.27   349.2 1816.79     388 1816.58   436.5  1816.7   446.1 1817.42
   455.8 1819.33  481.241826.991   484.7    1828   494.4 1829.83  515.451831.089
   590.9  1834.5   610.2  1835.7   639.2 1838.94   677.8 1844.16   697.1 1846.36
   706.7 1847.89   745.3 1858.32   803.2  1872.8   822.5 1878.21   841.8 1884.28
#Mann= 7 ,-1 , 0
       0     .12       0  210.65    .016       0   244.2     .12       0
   339.5    .045       0   446.1     .12       0  481.24    .016       0
  515.45     .12       0
Bank Sta=339.5,446.1
XS Rating Curve= 0 ,0
Exp/Cntr=0.3,0.1

Type RM Length L Ch R = 1 ,69503.8 ,401.8,406,410.2
XS GIS Cut Line= 3
      1804219.96      165372.846     1804194.363      164877.961
     1804169.875      164404.511
#Sta/Elev= 30
       0 1987.11    87.4 1948.21     136 1927.73   184.6 1903.88   223.5 1887.12
  253.31 1873.19  290.351857.467   310.9 1847.88   340.1    1832   359.5 1823.32
   369.2 1820.14     379 1818.39   388.7 1817.86     447 1816.49   485.8 1816.49
   495.6 1817.01  514.641823.751   524.6  1826.4  554.851829.451     573 1830.92
     602 1831.62   669.7 1829.46   708.4  1829.4   727.8 1830.18   747.1 1831.57
   785.8 1835.82   814.8 1841.52   843.8 1850.09   882.6 1862.97   969.6 1894.23
#Mann= 7 ,-1 , 0
       0     .12       0  253.31    .016       0  290.35     .12       0
   388.7    .045       0   495.6     .12       0  514.64    .016       0
  554.85     .12       0
Bank Sta=388.7,495.6
XS Rating Curve= 0 ,0
Exp/Cntr=0.3,0.1

Type RM Length L Ch R = 1 ,69097.7 ,604.7,613.9,623
XS GIS Cut Line= 3
     1804413.284       165407.59     1804589.249      165126.045
     1804611.124      164377.932
#Sta/Elev= 30
       0 1979.27     127 1935.66   136.7 1932.58   175.8 1922.32   263.7 1896.69
   312.5 1881.58   380.6 1862.57   409.8 1853.15  463.03 1833.89   497.2 1821.39
  504.341819.583     507 1818.91   516.7 1817.62   526.4 1817.05   545.8 1816.55
   594.4 1816.38   652.8 1816.54   662.5  1817.5   672.2 1819.84  680.371822.367
   691.6 1825.23   701.4 1826.29  716.931826.648   779.1 1828.73     818 1830.46
   895.8 1832.32   905.5 1833.73   915.2 1837.11  1022.1 1892.67  1080.4 1921.82
#Mann= 7 ,-1 , 0
       0     .12       0  463.03    .016       0  504.34     .04       0
   526.4    .045       0   652.8     .12       0  680.37    .016       0
  716.93     .12       0
Bank Sta=526.4,652.8
XS Rating Curve= 0 ,0
Exp/Cntr=0.3,0.1

Type RM Length L Ch R = 1 ,68483.9 ,880.8,904.3,927.8
XS GIS Cut Line= 4
     1804612.818      165483.587     1804957.863      165252.285
     1805177.791      164537.503     1805112.814      164324.007
#Sta/Elev= 30
       0 1948.19   125.6 1913.69   183.6 1901.98   289.8 1883.11   376.8  1861.7
  425.69 1846.33   444.9  1840.9   471.11837.996  479.741837.308  529.871832.963
   572.8 1829.24   592.5 1828.58   671.2 1828.97     809  1832.1   887.7 1831.37
   956.6  1828.3   966.4 1825.91  987.651818.351     996 1816.47  1005.8 1816.38
  1074.7 1816.54  1084.5 1818.18    10911821.437 1126.041833.517  1143.6 1843.51
  1192.4 1874.09  1250.6  1907.7  1289.4 1927.27  1337.9 1948.35  1386.4  1973.1
#Mann= 9 ,-1 , 0
       0     .12       0  425.69    .016       0   471.1     .12       0
  479.74     .06       0  529.87     .12       0  987.65    .045       0
  1084.5     .12       0    1091    .016       0 1126.04     .12       0
#XS Ineff= 2 , 0
          812.78 1921.95
Permanent Ineff=
       F       F
Bank Sta=987.65,1084.5
XS Rating Curve= 0 ,0
Exp/Cntr=0.3,0.1

Type RM Length L Ch R = 1 ,67579.6 ,554.4,550.8,547.2
XS GIS Cut Line= 3
     1805245.499      165916.606     1805245.499      165636.462
     1806019.797      165063.571
#Sta/Elev= 30
       0 1906.73    38.6  1897.4   231.8 1855.55  257.761850.529   280.1    1847
   348.9 1839.92   378.4 1835.59  401.051833.516   447.2 1831.03     516 1820.94
  544.531820.653  624.871820.573   683.1 1819.79   742.1 1814.27   810.9    1814
   840.4 1814.15   850.2 1816.19   869.8 1825.65   889.5 1830.39  898.941833.569
     919  1842.2   948.5 1859.04     978 1874.12  1007.4 1885.57  1086.1 1913.21
 1140.831934.238 1174.761947.501    1204 1958.54  1233.5 1968.47  1243.3 1972.61
#Mann= 10 ,-1 , 0
       0     .12       0  257.76    .016       0  401.05     .12       0
  544.53     .06       0  624.87     .12       0   742.1    .045       0
   840.4    .016       0  898.94     .12       0 1140.83    .016       0
 1174.76     .12       0
Bank Sta=742.1,840.4
XS Rating Curve= 0 ,0
Exp/Cntr=0.3,0.1

Type RM Length L Ch R = 1 ,67028.7 ,479.5,472,464.5
XS GIS Cut Line= 2
     1805509.655      166123.593     1806140.894      165549.739
#Sta/Elev= 30
       0 1945.34    39.2 1928.31    58.8 1921.12    68.6 1918.15   127.5 1903.83
   156.9 1893.59   176.5 1885.16   264.8 1844.17  282.481835.104     304    1823
   313.8 1818.62  333.711812.206  337.761811.504   343.2 1810.56   362.8 1810.08
   460.9 1810.21   470.7  1811.8   500.1 1823.93   509.9 1826.44   519.7 1827.42
   578.5 1829.27  598.881830.929  647.251836.165   686.4 1839.15     706 1841.77
   725.6 1846.81   774.6 1861.78  812.421870.404   833.5    1876   853.1 1884.43
#Mann= 9 ,-1 , 0
       0     .12       0  282.48    .016       0  333.71     .12       0
  337.76     .08       0   343.2    .045       0   460.9     .12       0
  598.88    .016       0  647.25     .12       0  812.42    .016       0
Bank Sta=343.2,460.9
XS Rating Curve= 0 ,0
Exp/Cntr=0.3,0.1

Type RM Length L Ch R = 1 ,66556.7 ,483,477.1,471.3
XS GIS Cut Line= 2
     1805946.065      166449.815     1806418.804      165798.202
#Sta/Elev= 30
       0 1943.87    58.9 1919.92   147.3  1886.1   166.9 1877.34     216 1852.72
  233.781844.198   245.4 1838.52   255.2 1832.61   265.1 1824.62   274.9 1816.23
   284.7 1811.71   294.5 1810.26   304.3 1810.08  395.251810.299   402.5 1810.78
   412.3 1812.85   441.8 1823.34   451.6 1825.52   461.4 1826.28   559.6 1828.36
   569.4 1829.16  598.921833.903  635.641838.306     648 1840.73   657.8 1843.17
   687.2  1851.4   716.7 1860.93   765.8  1878.3   775.6 1881.45     805 1889.63
#Mann= 6 ,-1 , 0
       0     .12       0  233.78    .016       0   294.5    .045       0
  395.25     .12       0  598.92    .016       0  635.64     .12       0
Bank Sta=294.5,395.25
XS Rating Curve= 0 ,0
Exp/Cntr=0.3,0.1

Type RM Length L Ch R = 1 ,66079.6 ,396.5,397.4,398.2
XS GIS Cut Line= 2
     1806401.017        166711.3     1806774.488      165981.931
#Sta/Elev= 30
       0 1928.17    19.5 1921.47    29.3 1918.61    58.5 1910.89   136.6 1888.62
   204.9 1867.88   263.4 1849.02   282.9 1843.06   312.2 1834.78  329.42 1830.69
   351.2 1824.96  366.351820.119   390.2 1812.46  399.821810.585   409.7 1810.12
   419.5 1810.08   526.8 1810.33   536.5 1811.35   546.3 1813.24  580.541821.197
   595.1 1824.79  619.651831.471   673.1 1846.14   682.9  1849.2   721.9 1863.26
   741.4 1869.51   770.6  1877.9   780.4 1881.35   799.9 1889.06   819.4 1895.14
#Mann= 7 ,-1 , 0
       0     .12       0  329.42    .016       0  366.35     .12       0
  399.82    .045       0   526.8     .12       0  580.54    .016       0
  619.65     .12       0
Bank Sta=399.82,526.8
XS Rating Curve= 0 ,0
Exp/Cntr=0.3,0.1

Type RM Length L Ch R = 1 ,65682.2 ,349.7,350,350.3
XS GIS Cut Line= 3
     1806728.425      166912.588     1806980.402      166447.401
     1807155.761      166123.661
#Sta/Elev= 30
       0 1931.22    68.6 1909.27   107.8 1897.25   244.9 1859.87   313.5 1841.96
   333.1 1837.66  397.311824.587   411.5 1821.59   421.3 1818.86  438.741812.903
   440.9 1812.18   450.7 1810.39   470.3 1810.08   606.6 1810.22   616.2  1811.2
   625.9 1814.32  630.271816.482   645.3 1823.37     655 1826.78   664.7 1829.29
  671.141830.605   713.1 1838.87   722.8 1840.95   732.5 1843.63   742.2 1847.03
   771.3 1858.41   790.6 1866.33   800.3 1870.81   858.5 1900.48   897.2 1919.85
#Mann= 7 ,-1 , 0
       0     .12       0  397.31    .016       0  438.74     .12       0
   450.7    .045       0   606.6     .12       0  630.27    .016       0
  671.14     .12       0
Bank Sta=450.7,606.6
XS Rating Curve= 0 ,0
Exp/Cntr=0.3,0.1

Type RM Length L Ch R = 1 ,65332.2 ,343.6,350,357.3
XS GIS Cut Line= 3
     1807016.926      167106.339     1807287.529      166615.243
     1807473.385       166277.95
#Sta/Elev= 30
       0 1942.55   108.2 1907.39   177.1 1886.61   196.7 1878.76   226.2 1863.49
  236.841860.747  249.741859.191   265.6 1857.68   295.1 1852.99   354.1 1837.78
   373.8 1833.56     423 1828.74  443.291824.743  476.161816.248   491.8 1811.83
   501.7  1810.3   511.5 1810.07  654.441810.759     657 1810.98   669.31817.541
   685.9 1826.77   695.5 1830.24  708.211833.369     734 1839.03   753.3  1844.7
   791.8 1860.07   820.7 1872.92   859.2 1886.17   916.9 1912.62   945.8 1922.95
#Mann= 9 ,-1 , 0
       0     .12       0  236.84     .06       0  249.74     .12       0
  443.29    .016       0  476.16     .12       0   501.7    .045       0
  654.44     .12       0   669.3    .016       0  708.21     .12       0
Bank Sta=501.7,654.44
XS Rating Curve= 0 ,0
Exp/Cntr=0.3,0.1

Type RM Length L Ch R = 1 ,64982.2 ,346.1,350,353
XS GIS Cut Line= 3
     1807222.771      167253.058     1807584.316      166799.199
     1807821.763      166515.794
#Sta/Elev= 30
       0  1946.4    29.5 1935.22    39.3 1932.05   216.4 1880.51   275.4 1862.72
  347.351841.697  387.191830.331   393.4 1828.74   403.2    1827   444.21823.283
   472.1 1820.16   481.9 1818.31  498.541814.002   511.4 1811.06   521.2 1810.14
   540.9 1810.08   658.1  1810.1   667.8 1811.07   677.6 1814.17  681.221816.193
     697 1825.03   706.8 1829.32  714.321832.142   735.9 1839.93   794.3 1860.11
   823.5 1870.69     843 1878.32   881.9  1891.1   920.8 1905.99     950 1916.38
#Mann= 9 ,-1 , 0
       0     .12       0  347.35     .06       0  387.19     .12       0
   444.2    .016       0  498.54     .12       0   521.2    .045       0
   658.1     .12       0  681.22    .016       0  714.32     .12       0
Bank Sta=521.2,658.1
XS Rating Curve= 0 ,0
Exp/Cntr=0.3,0.1

Type RM Length L Ch R = 1 ,64632.2 ,345.8,350,350.3
XS GIS Cut Line= 3
     1807459.172      167424.852     1807843.303      167034.319
     1808123.081      166749.878
#Sta/Elev= 30
       0 1943.72    19.6 1936.38    29.4 1933.15    58.7  1924.7   127.2 1902.91
   166.3 1889.63   244.6 1864.18   283.7 1850.32   303.2 1844.09   332.6 1836.64
   371.7 1827.85   381.5 1826.03  433.331820.277     450 1818.17  464.871814.289
   479.3 1810.69   489.1 1810.14   498.9 1810.08   606.2 1810.16   615.9 1811.64
   625.6 1815.96   635.4 1821.18   645.1 1825.32  657.641828.612   703.5 1839.58
     723 1844.81     830 1877.61   907.8 1903.14   927.3 1909.23   946.8 1915.94
#Mann= 6 ,-1 , 0
       0     .12       0  433.33    .016       0  464.87     .12       0
   479.3    .045       0   606.2    .016       0  657.64     .12       0
Bank Sta=479.3,606.2
XS Rating Curve= 0 ,0
Exp/Cntr=0.3,0.1

Type RM Length L Ch R = 1 ,64282.2 ,503,521.7,544.3
XS GIS Cut Line= 3
     1807686.367      167611.596     1808086.626      167285.829
     1808391.391      166981.063
#Sta/Elev= 30
       0 1943.42    48.7 1926.36   126.6 1899.69   175.3 1882.48   243.4 1857.98
   262.9 1851.56   311.6 1837.36   340.8 1829.28   350.5  1827.3   360.3 1825.94
  390.13 1822.73     409 1820.46   418.7 1818.64  432.341814.798   438.2 1813.04
   447.9 1810.76   457.6 1810.13   467.4 1810.08     565 1810.08   574.8 1810.15
   584.6 1810.89  636.191820.096     663 1824.61  682.561828.332   751.2  1842.4
     761 1844.51   770.8 1846.98   829.5 1863.79   868.7 1875.48   947.1 1897.58
#Mann= 7 ,-1 , 0
       0     .12       0  390.13    .016       0  432.34     .12       0
   447.9    .045       0   584.6     .12       0  636.19    .016       0
  682.56     .12       0
Bank Sta=447.9,584.6
XS Rating Curve= 0 ,0
Exp/Cntr=0.3,0.1

Type RM Length L Ch R = 1 ,63760.5 ,396.2,410,423.3
XS GIS Cut Line= 3
     1807839.459      167838.387     1808698.624      167678.128
     1808781.437      167746.413
#Sta/Elev= 30
       0 1930.84    19.6 1925.12    68.7 1909.64   166.9 1880.38   265.1 1846.75
   304.4 1834.02   324.1  1828.3  344.461823.738   363.3 1820.43  380.891815.973
   402.6 1810.87   412.4 1810.16   432.1 1810.08   540.1 1810.16  637.841814.242
   677.6 1814.45   687.4 1814.76   697.2 1815.85  738.471825.903   756.1 1830.05
  769.021832.104  832.531840.009   854.3 1842.74   864.2 1844.82     874 1847.48
  886.991852.996   893.5 1855.54   903.3 1858.44   942.3 1868.46   981.3 1879.22
#Mann= 10 ,-1 , 0
       0     .12       0  344.46    .016       0  380.89     .12       0
   412.4    .045       0   540.1     .08       0  637.84     .12       0
  738.47    .016       0  769.02     .12       0  832.53    .016       0
  886.99     .12       0
Bank Sta=412.4,540.1
XS Rating Curve= 0 ,0
Exp/Cntr=0.3,0.1

Type RM Length L Ch R = 1 ,63350.5 ,393.5,408.2,423.3
XS GIS Cut Line= 2
     1807874.304      168065.819     1808702.913       168210.08
#Sta/Elev= 30
       0 1911.13    29.3    1898    39.1 1894.14    58.7 1887.34    68.5  1884.4
    78.2 1882.09     176 1863.19   244.5 1848.46   264.1 1844.58   332.5 1832.77
   361.9 1828.76   371.6 1827.12  411.951818.984  438.981814.615  466.931810.958
   469.4 1810.64   479.2 1810.12     489 1810.08   586.8 1810.23   596.6 1812.32
   606.4  1817.1   616.1 1823.33  630.12 1833.11   635.7 1837.01   645.5 1842.85
   655.3 1847.09  661.141849.149   694.4  1861.1   772.6 1891.28   841.1 1915.43
#Mann= 8 ,-1 , 0
       0     .12       0  411.95    .016       0  438.98     .12       0
  466.93     .08       0   469.4    .045       0   586.8     .12       0
  630.12    .016       0  661.14     .12       0
Bank Sta=469.4,586.8
XS Rating Curve= 0 ,0
Exp/Cntr=0.3,0.1

Type RM Length L Ch R = 1 ,62942.3 ,508.7,528.9,549
XS GIS Cut Line= 2
      1807824.43      168265.556     1808543.249      168722.788
#Sta/Elev= 30
       0 1906.98      49 1888.55    78.3 1878.51   127.3 1864.22     186 1850.31
   215.4 1844.55     235 1841.22   264.4 1836.71   313.4 1830.06   352.5 1826.34
  406.371822.357   421.1 1821.08   430.8 1819.64  445.151816.363   460.2 1812.46
  471.561810.331   479.8  1809.7   489.6 1809.68   577.7  1809.7   587.5 1811.05
   597.3 1815.62   616.9 1830.98   626.7 1837.64   636.5 1843.05   646.3 1847.88
   665.9 1856.97     705 1872.54   734.4 1883.71   793.2 1904.63   851.9  1924.2
#Mann= 6 ,-1 , 0
       0     .12       0  406.37    .016       0  445.15     .12       0
  471.56    .045       0   577.7    .016       0   646.3     .12       0
Bank Sta=471.56,577.7
XS Rating Curve= 0 ,0
Exp/Cntr=0.3,0.1

Type RM Length L Ch R = 1 ,62413.4 ,421.6,441.1,460.6
XS GIS Cut Line= 3
     1807660.454      168444.211     1807975.534      169065.281
     1807981.948      169220.829
#Sta/Elev= 30
       0 1892.82      49 1879.21    68.7 1874.72    98.1 1866.41   127.5 1859.14
   176.6 1848.37   225.6 1838.92  246.42 1833.99   264.8 1829.05  284.511820.852
   304.1 1812.72   313.9 1810.17   333.5 1809.18   382.5 1809.31   402.2 1810.11
     412 1811.29   441.4 1816.59  480.231821.238   510.1  1824.1   559.1 1823.87
  573.021824.412  591.381825.333   608.1 1826.65     618 1828.78  631.291833.814
   657.2 1844.34   676.8 1851.23  747.921872.853  779.741882.389   852.1 1904.76
#Mann= 11 ,-1 , 0
       0     .12       0  246.42    .016       0  284.51     .12       0
   313.9    .045       0   402.2     .12       0  480.23     .06       0
  573.02     .12       0  591.38    .016       0  631.29     .12       0
  747.92    .016       0  779.74     .12       0
Bank Sta=313.9,402.2
XS Rating Curve= 0 ,0
Exp/Cntr=0.3,0.1

Type RM Length L Ch R = 1 ,61972.3 ,415.9,412.7,409.4
XS GIS Cut Line= 2
     1807447.029      168466.188     1807409.309      169269.926
#Sta/Elev= 30
       0 1902.15    39.2  1889.7    78.5  1877.9    98.1 1872.46   137.4 1862.63
     157 1857.34   196.2 1846.12   225.7 1837.89   235.5 1834.79  251.421829.333
   255.1 1828.09   264.9 1825.32  281.131821.792   304.2 1817.06     314 1815.28
   323.8  1813.8   353.2  1810.5   363.1  1809.6   372.9 1809.19   480.8  1809.1
   500.4 1809.31   510.2 1810.43   520.1  1813.1   559.3 1826.53   569.1 1829.98
     628 1851.75   667.2 1866.93   677.1 1870.53   775.2 1903.29   804.6  1913.6
#Mann= 5 ,-1 , 0
       0     .12       0  251.42    .016       0  281.13     .12       0
   372.9    .045       0   500.4     .12       0
Bank Sta=372.9,500.4
XS Rating Curve= 0 ,0
Exp/Cntr=0.3,0.1

Type RM Length L Ch R = 1 ,61559.6 ,431.9,423.9,415.8
XS GIS Cut Line= 2
     1806994.252      168447.415     1807026.302      169259.842
#Sta/Elev= 30
       0 1891.79   137.1 1855.08   186.1 1840.89   195.9 1838.42   235.1  1829.6
   244.9 1827.89   254.7 1826.64   264.5 1825.81   274.3  1825.4   284.1 1825.33
   323.3 1826.14   333.1 1825.82  337.651825.295   342.9 1824.69   352.6 1822.58
   362.4 1820.78  369.771820.517     382 1820.23   391.8 1818.53   411.4 1811.89
   421.2 1809.72     431 1809.08   519.2 1809.18     529 1810.41   538.8 1813.35
   568.2 1824.07   607.4 1838.72   685.7 1868.57   764.1  1899.4   813.1 1919.25
#Mann= 5 ,-1 , 0
       0     .12       0  337.65    .016       0  369.77     .12       0
   421.2    .045       0     529     .12       0
Bank Sta=421.2,529
XS Rating Curve= 0 ,0
Exp/Cntr=0.3,0.1

Type RM Length L Ch R = 1 ,61135.7 ,451.9,439.8,427.8
XS GIS Cut Line= 3
     1806438.423      168556.773     1806529.203      168690.106
       1806685.9        169305.7
#Sta/Elev= 30
       0 1898.96      38 1889.82    66.4 1880.96    85.4 1875.63   104.4 1871.33
   132.8 1866.46   142.3 1864.51   151.8 1861.57   161.3 1857.59   190.6  1843.3
   200.4 1838.94   210.2 1835.27   219.9 1832.65  293.621818.497   307.9 1815.77
  318.691812.858   327.4 1810.46   337.2 1809.28     347 1809.08   444.7 1809.32
   454.5 1810.24   464.3 1811.97   513.1 1821.71   522.9 1824.56   581.5 1847.97
   610.8 1858.43   669.5 1876.09   737.9 1898.07     777  1912.2   796.5 1919.67
#Mann= 5 ,-1 , 0
       0     .12       0  293.62    .016       0  318.69     .08       0
   337.2    .045       0   444.7     .12       0
Bank Sta=337.2,444.7
XS Rating Curve= 0 ,0
Exp/Cntr=0.3,0.1

Type RM Length L Ch R = 1 ,60695.8 ,421.7,418.3,414.8
XS GIS Cut Line= 2
     1806008.399      168806.702     1806415.244      169439.572
#Sta/Elev= 30
       0 1896.84    39.1 1887.44    48.8 1884.47    58.6 1880.79    97.7 1864.75
   107.5 1860.98   117.2 1857.74   136.8 1854.19   146.6 1851.77   195.4  1836.6
   205.2 1834.09  243.761825.704     254 1823.32   263.8 1819.44   273.6 1814.05
   283.4 1810.32  289.941809.518   293.1 1809.13   302.9 1809.08   390.8 1809.12
  401.291809.664   410.4 1810.78   459.2 1819.25   488.6 1823.52   498.3 1825.76
   508.1 1828.95   547.2 1843.82   615.6 1871.29   654.6 1886.26   752.4 1926.04
#Mann= 4 ,-1 , 0
       0     .12       0  243.76    .016       0  289.94    .045       0
  401.29     .12       0
Bank Sta=289.94,401.29
XS Rating Curve= 0 ,0
Exp/Cntr=0.3,0.1

Type RM Length L Ch R = 1 ,60277.5 ,491.5,477.3,462.9
XS GIS Cut Line= 2
     1805644.223      169065.287     1806089.441      169634.364
#Sta/Elev= 30
       0 1908.19    48.8 1888.33    58.6 1884.64    97.6 1871.86   136.7  1858.5
     205 1833.27  219.271828.405   234.3 1823.38   244.1 1819.47   253.9 1814.68
  263.06 1810.94   273.4 1809.25   283.2 1809.08   380.8 1809.14   390.6 1809.69
   400.3 1811.18   439.4 1818.55   458.9 1822.68   468.7 1825.31   546.8 1848.54
   585.8 1859.76   624.9 1872.71   644.4 1878.56   654.2 1880.98     664 1882.86
   673.7 1884.23   693.2 1886.05     703 1887.72   712.8 1890.62   722.5 1894.53
#Mann= 5 ,-1 , 0
       0     .12       0  219.27    .016       0  263.06     .12       0
   273.4    .045       0   380.8     .12       0
Bank Sta=273.4,380.8
XS Rating Curve= 0 ,0
Exp/Cntr=0.3,0.1

Type RM Length L Ch R = 1 ,59800.2 ,457.1,437.6,417.7
XS GIS Cut Line= 2
      1805215.41      169488.267     1805873.731      169872.288
#Sta/Elev= 30
       0 1898.37    29.3 1888.58    58.6 1881.17    87.9 1875.45    97.7 1873.03
   107.5 1870.41   156.3 1855.49   195.4 1844.71   205.2 1842.17   224.7 1837.56
  282.741824.902   293.1 1821.69   312.7 1811.62  322.211809.316   325.91809.202
   332.2 1809.08   429.9  1809.2   439.7 1810.11   478.8 1816.98   508.1 1821.74
   537.4 1827.03   547.2 1829.25     557 1831.94   586.3 1841.42   615.6 1850.08
   635.1 1856.18   693.7 1875.79   742.6 1891.11   752.4 1894.42   762.1 1897.99
#Mann= 5 ,-1 , 0
       0     .12       0  282.74    .016       0  322.21     .12       0
   325.9    .045       0   429.9     .12       0
Bank Sta=325.9,429.9
XS Rating Curve= 0 ,0
Exp/Cntr=0.3,0.1

Type RM Length L Ch R = 1 ,59362.6 ,511.8,500.9,489.9
XS GIS Cut Line= 2
     1804847.966      170099.863      1805811.98      170106.377
#Sta/Elev= 30
       0 1892.93      59 1873.92    98.4 1863.36     118 1859.14   147.6  1854.6
   177.1 1848.68   206.6 1844.35   255.8 1838.33   314.8 1832.68   383.6    1828
  525.961820.193     541 1819.87   550.9 1817.03   560.7 1812.06  564.651811.027
   570.6 1809.47   580.4 1809.07   659.1 1809.12   668.9 1809.75   678.8 1811.69
   708.3 1820.89   718.1 1823.08     728  1823.4   757.5 1821.29   767.3 1821.98
   777.1 1823.91   806.6 1832.48   826.3 1840.86   885.3 1869.52     964 1910.56
#Mann= 5 ,-1 , 0
       0     .12       0  525.96    .016       0  564.65     .04       0
   580.4    .045       0   659.1     .12       0
Bank Sta=580.4,659.1
XS Rating Curve= 0 ,0
Exp/Cntr=0.3,0.1

Type RM Length L Ch R = 1 ,58861.7 ,633.7,600.2,565.3
XS GIS Cut Line= 3
     1804765.279      170693.449     1805063.925      170736.113
     1805872.783      170499.678
#Sta/Elev= 30
       0 1934.73    38.9 1922.94   136.2 1891.18   214.1 1867.35   272.5 1850.93
   331.1 1835.79  362.371826.497   370.3 1824.96   380.1 1824.26   468.3 1822.51
   546.6 1822.48   605.4 1823.05  704.681819.121     723  1818.9   732.8 1818.14
  735.311817.133   752.4 1810.31   762.2 1809.08   850.4 1809.16   860.2 1809.98
   889.6 1819.39   899.4 1821.71   938.6 1827.75   948.4 1830.14   977.8 1841.07
   997.4 1847.64  1036.6 1858.82  1075.8 1871.88  1085.6 1874.75  1144.4 1889.82
#Mann= 6 ,-1 , 0
       0     .12       0  362.37     .06       0  704.68    .016       0
  735.31     .12       0   762.2    .045       0   850.4     .12       0
Bank Sta=762.2,850.4
XS Rating Curve= 0 ,0
Exp/Cntr=0.3,0.1

Type RM Length L Ch R = 1 ,58261.5 ,786.9,751.5,716.6
XS GIS Cut Line= 3
     1805729.107       171663.14     1805640.465      171409.031
      1805996.68      170579.087
#Sta/Elev= 30
       0 1964.89    86.5  1941.6   105.7 1935.01   115.3  1930.7   230.7 1867.49
  268.581843.568   278.9 1838.31   288.8 1834.54  302.011831.024     328 1824.84
   337.8 1823.94  415.671823.964   445.8 1823.43   455.6 1821.45  480.921812.048
   494.9 1809.14   583.3 1809.07   593.1 1809.25   602.9 1810.82   642.2 1821.94
   661.8 1825.37   779.6 1829.27   887.6 1830.22   956.3 1836.42   995.6 1838.01
  1015.2 1841.75  1044.7 1850.05  1083.9 1857.41    1133 1868.87  1172.3 1875.58
#Mann= 7 ,-1 , 0
       0     .12       0  268.58    .016       0  302.01     .12       0
  415.67    .016       0  480.92     .12       0   494.9    .045       0
   593.1     .12       0
#XS Ineff= 2 , 0
          383.95 1945.12
Permanent Ineff=
       F       F
Bank Sta=494.9,593.1
XS Rating Curve= 0 ,0
Exp/Cntr=0.3,0.1

Type RM Length L Ch R = 1 ,57510   ,508.6,524.1,539.6
XS GIS Cut Line= 3
     1806555.707      171313.378     1806456.437      171005.385
      1806166.38      170526.792
#Sta/Elev= 30
       0 1948.44    39.2 1930.76    58.8 1923.76   117.7 1907.02   215.7 1877.51
   264.8 1864.38     304 1852.87   313.8 1850.25   343.2 1845.05   372.7 1838.88
   382.5 1835.97  402.521826.764     412 1823.24   431.6 1820.54   441.4 1818.37
     461 1810.45   470.9 1808.37   480.7 1807.79   578.9 1808.43   588.7 1809.95
   618.1 1820.11     628 1821.99   667.2 1822.37   706.5 1824.67   716.3 1825.91
   726.1 1828.33   775.2 1845.71   824.3 1861.91     844  1869.6   883.2  1886.3
#Mann= 4 ,-1 , 0
       0     .12       0  402.52    .016       0   470.9    .045       0
   578.9     .12       0
Bank Sta=470.9,578.9
XS Rating Curve= 0 ,0
Exp/Cntr=0.3,0.1

Type RM Length L Ch R = 1 ,56985.9 ,645.9,667,688.1
XS GIS Cut Line= 2
     1806859.567      171166.452     1806749.092      170337.885
#Sta/Elev= 30
       0 1922.22     9.8 1917.58    39.3 1900.45      59 1889.98    68.8  1885.2
    78.7 1881.67    98.3 1878.21   127.8 1875.63   137.7 1873.96   186.8 1859.95
   245.8 1846.13   285.2 1838.27   324.5 1829.39     354 1824.93   403.2 1821.16
   501.5 1822.01   511.4  1821.4  520.471819.669     531 1817.06  565.391812.094
   580.2  1808.9  595.13 1807.69   599.9 1807.57   658.9 1807.83   668.7 1809.18
   678.6 1812.44   688.4 1817.15   767.1 1859.39   786.7 1870.66   835.9 1903.13
#Mann= 5 ,-1 , 0
       0     .12       0  520.47    .016       0  565.39     .12       0
  595.13    .045       0   658.9     .12       0
Bank Sta=595.13,658.9
XS Rating Curve= 0 ,0
Exp/Cntr=0.3,0.1

Type RM Length L Ch R = 1 ,56318.9 ,434.8,436.7,438.7
XS GIS Cut Line= 2
     1807162.525      171176.503     1807500.937      170447.165
#Sta/Elev= 30
       0 1908.78    58.8 1888.43    78.4 1881.92   215.7 1844.04   235.3 1839.51
   294.2  1827.4   333.4 1819.92  349.211817.311     353 1816.75  378.171814.691
   382.4 1814.19     402 1808.88   411.8 1807.66   421.6 1807.58   500.1 1807.64
   509.9 1807.97   519.7 1809.23   529.5  1811.4   539.3 1813.98   549.1 1816.87
   588.3 1829.49   598.1 1831.21   637.3 1836.74   647.1 1838.86     657 1841.73
   715.8 1861.92   745.2 1875.02     755 1878.32   784.4 1885.83     804  1891.8
#Mann= 5 ,-1 , 0
       0     .12       0  349.21    .016       0  378.17     .12       0
   411.8    .045       0   509.9     .12       0
Bank Sta=411.8,509.9
XS Rating Curve= 0 ,0
Exp/Cntr=0.3,0.1

Type RM Length L Ch R = 1 ,55882.2 ,310.1,322.1,333.1
XS GIS Cut Line= 3
     1807547.516      171326.139      1807734.24      170968.252
     1807904.077       170642.73
#Sta/Elev= 30
       0 1895.42    19.2 1889.65    38.4  1884.6   105.7  1867.7   192.2 1846.44
  299.791824.009   307.6 1822.74   326.8 1820.57   336.4  1816.9     346 1811.71
   355.6 1808.42   365.2 1807.39   384.4 1807.21     452 1807.53   461.6 1808.07
   471.3 1809.47     510 1819.58   519.6 1821.65   529.3 1823.34   538.9 1824.62
   548.6 1825.53   577.6 1827.19   587.2 1829.14   596.9 1832.33   616.2 1839.94
   635.6 1846.81   654.9 1854.33   664.6 1857.74   722.5 1876.38   770.8 1893.19
#Mann= 4 ,-1 , 0
       0     .12       0  299.79    .016       0   365.2    .045       0
     452     .12       0
Bank Sta=365.2,452
XS Rating Curve= 0 ,0
Exp/Cntr=0.3,0.1

Type RM Length L Ch R = 1 ,55560.1 ,384.5,392.4,400.5
XS GIS Cut Line= 3
     1807669.989      171447.983     1807985.044      171161.777
     1808243.208      170896.992
#Sta/Elev= 30
       0 1897.78    67.7 1881.52   106.4 1871.34   125.8 1866.83   145.1 1863.06
   270.9 1840.66   328.9 1828.73  349.821823.714   357.9 1822.04   377.3 1820.03
     387 1818.47  402.631813.753     416 1809.24   425.6 1806.98   435.4 1806.16
     523 1808.62   532.7  1809.2   542.4 1810.96   552.2 1814.74   571.6 1823.33
   581.4 1825.91   591.1 1827.34   620.3 1830.53   649.5 1834.52   668.9 1838.12
   688.4 1843.24   707.9 1849.45   756.5 1868.48   766.3 1872.78   795.5 1887.32
#Mann= 5 ,-1 , 0
       0     .12       0  349.82    .016       0  402.63     .12       0
   425.6    .045       0     523     .12       0
Bank Sta=425.6,523
XS Rating Curve= 0 ,0
Exp/Cntr=0.3,0.1

Type RM Length L Ch R = 1 ,55167.7 ,411.9,417.2,423.6
XS GIS Cut Line= 3
     1807828.718      171712.291     1808200.295      171479.375
     1808537.167      171257.722
#Sta/Elev= 30
       0 1922.41    68.2 1895.21   116.9 1877.26   136.4 1871.34   204.6 1852.75
  287.561828.445   302.1 1825.43  314.481823.856  344.691820.291   360.6 1819.32
  371.96  1817.5   380.1  1815.1   399.6 1807.18   409.3 1804.76  414.211804.391
   428.8 1803.98   497.6 1804.09   507.4 1804.85   517.2 1807.66   536.9 1816.99
   546.7 1820.67   556.6  1822.8   654.9 1830.26   664.8 1831.87   723.8 1845.33
   743.4 1850.46   753.3 1853.64   802.4 1871.11     832 1880.52   841.8  1884.8
#Mann= 7 ,-1 , 0
       0     .12       0  287.56     .06       0  314.48     .12       0
  344.69    .016       0  371.96     .12       0  414.21    .045       0
   497.6     .12       0
Bank Sta=414.21,497.6
XS Rating Curve= 0 ,0
Exp/Cntr=0.3,0.1

Type RM Length L Ch R = 1 ,54750.5 ,494.6,504.6,514
XS GIS Cut Line= 3
     1807964.409      172041.464      1808374.61      171855.604
     1808764.787      171686.141
#Sta/Elev= 30
       0 1920.44    19.6 1912.29    58.7 1894.14   127.3 1867.66   137.1 1865.52
   156.6  1862.7   176.2 1858.53   195.8 1853.38   244.8  1838.4   264.3 1833.22
   303.5 1824.22  342.341816.916     372 1813.49  376.781811.812   391.6 1805.98
   401.4 1804.08     489 1803.96   498.7 1804.65   508.4 1807.55     518 1812.02
   527.7 1815.73   537.4 1817.42     634 1819.11   653.4 1819.85     663 1821.15
   682.4 1826.44     750 1848.37   808.1 1866.13   846.7 1881.34   875.7 1891.76
#Mann= 5 ,-1 , 0
       0     .12       0  342.34    .016       0  376.78     .12       0
   401.4    .045       0     489     .12       0
Bank Sta=401.4,489
XS Rating Curve= 0 ,0
Exp/Cntr=0.3,0.1

Type RM Length L Ch R = 1 ,54245.9 ,393,396,399.1
XS GIS Cut Line= 3
     1807955.674      172319.203     1808157.241      172372.745
     1808897.825      172252.185
#Sta/Elev= 30
       0 1926.24    85.3 1897.27   123.2 1885.02   170.6 1871.14   276.8 1838.82
   286.5 1835.81     306 1828.86   315.8 1826.13   325.5 1824.66  343.761823.312
  368.631821.911   422.9 1820.41  487.651820.931   539.9 1821.18  549.751820.491
   569.1 1815.03   588.6 1812.22  591.291811.338   608.1 1805.65   617.8 1804.14
   705.5 1803.97   715.3 1804.11     725 1806.24   734.8 1810.44   744.5  1813.8
   754.2 1816.42     764 1820.43   783.5 1831.48   793.2 1835.82   958.9 1895.49
#Mann= 8 ,-1 , 0
       0     .12       0  343.76     .08       0  368.63     .06       0
  487.65     .12       0  549.75    .016       0  591.29     .12       0
   617.8    .045       0   715.3     .12       0
#XS Ineff= 2 , 0
          523.46  1879.8
Permanent Ineff=
       F       F
Bank Sta=617.8,715.3
XS Rating Curve= 0 ,0
Exp/Cntr=0.3,0.1

Type RM Length L Ch R = 1 ,53849.8 ,370.5,364.3,357.9
XS GIS Cut Line= 3
     1807913.919      172611.127     1808115.575       172732.12
     1808983.987      172662.248
#Sta/Elev= 30
       0 1893.23    58.8 1877.63   107.8 1865.37   156.8 1855.52   235.2 1838.93
  271.681834.037   342.8 1826.04     431 1824.38   450.5 1823.39   509.3 1818.88
   548.4 1818.42   665.9 1819.73   675.7 1819.43  678.371818.863   685.5 1817.35
   695.2  1813.3     705  1810.5   718.6 1808.25   734.4 1804.56     754 1803.98
   822.5 1804.04   832.3  1805.1   842.1 1809.56   861.7 1823.38   871.4 1829.02
   881.2 1833.24   920.4  1846.3   959.6 1860.54  1018.3 1883.69  1106.4 1919.39
#Mann= 6 ,-1 , 0
       0     .12       0  271.68     .06       0  678.37    .016       0
   718.6     .12       0   734.4    .045       0   832.3     .12       0
Bank Sta=734.4,832.3
XS Rating Curve= 0 ,0
Exp/Cntr=0.3,0.1

Type RM Length L Ch R = 1 ,53485.5 ,302.7,298.6,294.1
XS GIS Cut Line= 3
     1807806.966      173261.165     1808084.325       173200.87
     1809047.103      172957.744
#Sta/Elev= 30
       0 1921.21    39.2 1903.04    58.7 1895.71    97.9 1882.58     137 1865.46
   146.8 1861.87   166.4 1856.98  258.671841.192  292.791835.395  323.131830.182
   352.7 1826.26   382.2 1824.35   411.6 1823.04  486.141821.601  505.181821.354
     569 1820.99  643.531818.606  675.651817.302  744.381814.411   824.6 1808.78
  838.941805.856   844.2 1804.75   854.1 1804.04   932.7 1803.94   942.6 1804.73
  946.861805.921  1011.4 1829.67  1060.5  1846.4  1139.2 1879.73  1276.8 1933.85
#Mann= 12 ,-1 , 0
       0     .12       0  258.67     .08       0  292.79     .12       0
  323.13     .06       0  486.14     .08       0  505.18     .06       0
  643.53     .12       0  675.65     .06       0  744.38    .016       0
  838.94     .08       0   844.2    .045       0  946.86     .12       0
Bank Sta=844.2,946.86
XS Rating Curve= 0 ,0
Exp/Cntr=0.3,0.1

Type RM Length L Ch R = 1 ,53186.9 ,238.9,243.1,261.1
XS GIS Cut Line= 3
     1807836.645      173665.976     1809134.388      173192.885
     1809296.638      173144.302
#Sta/Elev= 30
       0 1880.14    68.6 1872.39  107.291862.587   127.4  1858.3  166.181864.618
  185.651865.135   216.91861.226   264.5 1852.45   293.9 1848.87   489.8 1835.12
   568.2 1835.55   617.2 1832.61   744.5 1816.58   782.71814.632  810.731813.188
   832.7 1812.45  849.911809.152   862.1 1805.73   881.7 1803.98     960 1803.97
   979.6 1805.96    1058 1820.17    1156 1827.73  1224.5 1845.77  1283.3 1864.41
  1322.5 1871.18  1381.3 1875.75  1484.8 1880.69 1539.241880.883  1550.6 1880.74
#Mann= 11 ,-1 , 0
       0     .06       0  107.29     .08       0  166.18    .016       0
  185.65     .08       0   216.9     .06       0   782.7     .08       0
  810.73    .016       0  849.91     .12       0   862.1    .045       0
   979.6     .12       0 1539.24     .08       0
Bank Sta=862.1,979.6
XS Rating Curve= 0 ,0
Exp/Cntr=0.3,0.1

Type RM Length L Ch R = 1 ,52943.8 ,874.7,817.5,746.9
XS GIS Cut Line= 3
     1807927.791      173904.691     1809212.513      173401.219
     1809571.871      173293.614
#Sta/Elev= 30
       0 1843.62   27.181842.554   53.651841.769   96.581840.233  180.681836.821
   303.4 1831.59  377.921829.174  440.971827.172  448.381826.938   516.51824.796
  567.061824.264     734 1823.68   753.5 1821.38   802.5 1812.35  819.261810.388
   861.2 1809.99  872.241808.591   890.5 1804.73   910.1 1803.98  1017.8 1803.98
  1037.3 1804.97  1056.9 1807.59    1096 1814.43  1105.8 1815.15  1213.5 1820.57
 1378.25 1827.36 1417.191827.777 1482.961829.146  1687.6 1832.72    1755 1833.24
#Mann= 17 ,-1 , 0
       0     .12       0   27.18     .06       0   53.65     .12       0
   96.58     .06       0  180.68     .12       0  377.92     .06       0
  440.97     .12       0  448.38     .06       0   516.5     .08       0
  567.06     .06       0  819.26    .016       0  872.24     .12       0
   890.5    .045       0  1037.3     .12       0 1378.25     .08       0
 1417.19     .12       0 1482.96     .06       0
Bank Sta=890.5,1037.3
XS Rating Curve= 0 ,0
Exp/Cntr=0.3,0.1

Type RM Length L Ch R = 1 ,52126.3 ,556.1,552.8,549.5
XS GIS Cut Line= 2
     1809690.227      173815.453     1809596.477      173280.731
#Sta/Elev= 30
       0 1858.93    19.4 1853.59    58.2  1843.2    77.6 1838.25    96.9 1833.61
   116.3 1829.26   155.1 1821.36   174.5 1817.63  184.02 1816.04   193.9 1814.89
   213.3 1813.49  217.441812.837     223 1811.96     252 1805.59   261.7 1804.35
   271.4 1803.98   387.8 1803.98   397.5 1804.38   407.2  1806.3   416.8 1809.53
   426.6  1813.2   436.2 1816.52   445.9 1818.79   455.6 1819.81     475 1820.71
  478.361821.022   484.7 1821.61   494.4 1823.24   504.1 1825.41   542.9 1834.76
#Mann= 6 ,-1 , 0
       0     .12       0  184.02    .016       0  217.44     .12       0
   261.7    .045       0   387.8     .12       0  478.36     .06       0
Bank Sta=261.7,387.8
XS Rating Curve= 0 ,0
Exp/Cntr=0.3,0.1

Type RM Length L Ch R = 1 ,51573.5 ,543,551.5,560
XS GIS Cut Line= 2
     1810273.561      173780.731     1810096.477      173114.064
#Sta/Elev= 30
       0 1899.21    58.3 1875.99    87.4 1863.12     136 1843.16   174.9 1828.56
  186.251824.902   194.3 1823.06   213.7  1820.3  225.881816.014   242.9 1808.27
   252.6 1805.19   262.3 1803.89     272 1803.86   378.9 1803.99   388.6  1804.8
   398.3 1806.88   427.5 1815.23   437.2 1817.62   446.9 1819.45   456.6 1820.51
     476  1821.3   495.5 1821.48   544.1 1820.67   582.9  1820.6   602.4 1820.79
   612.1 1821.56   621.8  1823.7   631.5 1826.99  657.621837.111   689.8  1848.3
#Mann= 6 ,-1 , 0
       0     .12       0  186.25    .016       0  225.88     .12       0
   262.3    .045       0   378.9     .12       0  657.62     .06       0
Bank Sta=262.3,378.9
XS Rating Curve= 0 ,0
Exp/Cntr=0.3,0.1

Type RM Length L Ch R = 1 ,51022   ,470.8,498.3,525.7
XS GIS Cut Line= 2
     1810745.783      173808.509     1810708.127      172712.271
#Sta/Elev= 30
       0 1936.38      49 1925.97    97.9  1909.5   127.3 1896.43   176.3 1870.46
   225.2 1846.42  247.171837.742   264.4 1834.52   274.2 1830.46   303.6 1810.06
   313.4 1806.79   323.2 1805.95   440.7 1803.69   450.5 1803.94   460.3 1805.22
   489.7 1813.43   509.3  1815.7   538.6 1816.34  582.021813.034  601.061811.872
     617 1812.16   626.8 1813.94  691.361832.251   714.9 1835.48   763.9 1837.26
  998.341840.231  1018.5  1840.3 1049.281844.065 1079.53 1848.61  1096.9 1850.83
#Mann= 10 ,-1 , 0
       0     .12       0  247.17    .016       0   323.2    .045       0
   450.5     .12       0  582.02     .06       0  601.06     .12       0
  691.36     .06       0  998.34     .08       0 1049.28     .06       0
 1079.53     .12       0
Bank Sta=323.2,450.5
XS Rating Curve= 0 ,0
Exp/Cntr=0.3,0.1

Type RM Length L Ch R = 1 ,50523.8 ,433.7,457.8,481.9
XS GIS Cut Line= 3
     1810856.894       173857.12     1811346.477      173266.842
     1811575.343      173192.865
#Sta/Elev= 30
       0 1914.09    29.5 1907.12    78.7 1894.41   108.2 1885.88   147.5 1873.04
   186.8  1861.7   275.3 1837.46   324.4 1825.39   344.1 1821.82     354    1821
   383.4 1820.46  412.711820.925   422.8 1821.12   432.6 1820.53   442.4 1818.37
   452.3 1813.52   462.1 1807.92   471.9 1805.53   481.8 1804.77   521.1 1803.58
   629.2 1803.62   639.1    1804   648.9  1805.2   678.4 1811.05   707.9 1817.95
   805.4 1842.26   853.5 1851.72     892 1860.77   920.8 1866.52  1007.4  1888.5
#Mann= 4 ,-1 , 0
       0     .12       0  412.71    .016       0   481.8    .045       0
   639.1     .12       0
Bank Sta=481.8,639.1
XS Rating Curve= 0 ,0
Exp/Cntr=0.3,0.1

Type RM Length L Ch R = 1 ,50066   ,364.9,369.2,373.5
XS GIS Cut Line= 2
      1810912.45       173919.62      1811776.04      173710.967
#Sta/Elev= 30
       0 1902.89    87.9    1879   214.8 1846.08   263.6 1831.86   283.1 1826.79
   292.9 1824.82   302.7 1823.41   322.2 1821.43   390.5 1815.46  426.42 1813.53
   439.3 1812.72   449.1 1811.18  463.261807.433   468.6 1805.93   478.4  1803.9
   488.2 1803.55   595.6 1803.65   605.3 1804.97   615.1 1808.75   644.4 1823.73
   654.1  1828.1   663.9 1831.32   693.2 1838.58   712.7 1844.51   722.5 1847.18
   761.5 1856.04     781 1860.89   800.6 1866.66   849.4 1881.74   888.4 1895.16
#Mann= 5 ,-1 , 0
       0     .12       0  426.42    .016       0  463.26     .12       0
   478.4    .045       0   605.3     .12       0
Bank Sta=478.4,605.3
XS Rating Curve= 0 ,0
Exp/Cntr=0.3,0.1

Type RM Length L Ch R = 1 ,49696.8 ,394.5,398.5,402.6
XS GIS Cut Line= 3
     1810948.383      174225.852     1811491.727      174158.534
     1811851.816       174113.92
#Sta/Elev= 30
       0  1899.8    68.4  1879.9   107.5 1868.88     176 1851.54   254.2 1830.68
   293.3 1821.29   312.9 1817.16   322.6 1815.35   332.4 1814.03     352  1812.3
   371.5 1811.25   400.8 1810.04  422.361808.632   430.2 1807.96  448.821804.432
   449.7 1804.26   459.5 1803.65   469.3 1803.58   586.7 1803.57   596.5 1804.07
   606.3 1805.96   635.8 1814.91   655.4 1821.36   694.6 1834.89     724 1844.68
   782.9 1862.66   822.1 1874.96   841.7 1881.46   871.1 1891.55   910.3 1905.53
#Mann= 5 ,-1 , 0
       0     .12       0  422.36    .016       0  448.82     .12       0
   449.7    .045       0   596.5     .12       0
Bank Sta=449.7,596.5
XS Rating Curve= 0 ,0
Exp/Cntr=0.3,0.1

Type RM Length L Ch R = 1 ,49298.2 ,353.5,356.6,360.3
XS GIS Cut Line= 3
     1810975.519      174564.835     1811518.749      174555.854
     1811862.178      174550.176
#Sta/Elev= 30
       0 1900.26    67.9 1880.49      97  1872.9   135.8  1864.3     194 1853.18
   213.4 1848.89   242.6 1841.76     262 1836.43   281.4 1830.36   300.8 1823.85
   320.2  1816.8   329.9 1813.78   339.6 1812.19   349.3 1811.75   397.8 1811.01
  436.031810.089   446.3 1809.19   465.7 1805.09  477.531803.783   485.1 1803.58
   602.2 1803.77     612 1805.45   621.8 1809.76   631.6 1815.29   641.4  1820.2
   651.2 1824.24   690.5 1838.79   729.8 1854.44   837.7 1902.82   886.8 1923.88
#Mann= 4 ,-1 , 0
       0     .12       0  436.03    .016       0  477.53    .045       0
   602.2     .12       0
Bank Sta=477.53,602.2
XS Rating Curve= 0 ,0
Exp/Cntr=0.3,0.1

Type RM Length L Ch R = 1 ,48941.6 ,405.8,409.3,412.3
XS GIS Cut Line= 3
     1810989.803      174877.043      1811525.49      174912.704
     1811850.164      174939.759
#Sta/Elev= 30
       0 1908.82    78.1 1882.03    87.8    1878   117.1 1864.33   126.9 1860.54
   136.7 1857.62   146.4 1855.53   156.2 1854.15   165.9 1853.45   195.2 1852.63
     205 1851.64   214.8 1849.84   224.5 1846.89   253.8 1834.93   302.6 1816.98
   312.4 1814.69   322.1 1813.73  413.071811.535   429.5 1810.54  445.51 1806.68
   458.8 1803.84   584.8 1803.54   594.4  1805.4   623.1 1821.96   632.7 1826.96
   642.3 1830.63   661.4 1835.47     671 1838.67   766.8 1881.04   862.7  1922.3
#Mann= 5 ,-1 , 0
       0     .12       0  413.07    .016       0  445.51     .12       0
   458.8    .045       0   584.8     .12       0
Bank Sta=458.8,584.8
XS Rating Curve= 0 ,0
Exp/Cntr=0.3,0.1

Type RM Length L Ch R = 1 ,48532.3 ,426.4,425.7,425
XS GIS Cut Line= 3
     1810987.873      175238.439     1811469.939      175316.323
     1811836.725      175375.581
#Sta/Elev= 30
       0 1916.54    19.5 1909.17    58.6 1894.97    97.7  1880.2     127  1867.5
   175.8 1844.71   185.6 1840.43   195.3 1837.17   205.1  1835.1   234.4 1830.01
   253.9 1826.17     293 1816.46   302.8 1814.44   312.5 1813.22  391.951805.729
   410.2 1804.07     420 1803.66   439.5 1803.58     547 1803.59   556.8 1804.14
   566.5  1806.4   605.6  1820.7   742.5 1861.06   762.1 1867.26   781.6 1874.34
   801.2 1882.04     811 1886.21   840.3  1899.5   850.1 1903.34   859.9 1906.52
#Mann= 4 ,-1 , 0
       0     .12       0  391.95    .016       0     420    .045       0
     547     .12       0
Bank Sta=420,547
XS Rating Curve= 0 ,0
Exp/Cntr=0.3,0.1
