HEC-RAS study MIDFKRV2.prj: MIDFKRV2

--- MIDFKRV2.g01 (geometry) --- (continued)

Type RM Length L Ch R = 1 ,48106.6 ,460.4,466.3,472.2
XS GIS Cut Line= 3
     1810940.914      175670.458     1811425.871      175739.849
     1811805.065      175794.106
#Sta/Elev= 30
       0 1908.16      49 1887.91    78.4 1873.26    88.2 1869.83      98 1867.87
   107.8 1866.89   156.8 1864.47   166.6    1863   176.4 1860.21   186.2 1856.56
     245 1831.52   264.5 1823.78   284.1 1817.32   293.9 1814.59   303.7 1812.65
   313.5  1811.6   396.51806.799  418.181804.542   431.1 1803.57   548.8 1803.56
   558.6 1803.77   568.5 1805.16   597.9 1811.84   607.8 1814.39   617.6 1817.61
   686.3 1844.91   755.1 1867.72   804.2 1884.89   853.3 1903.42     873 1909.68
#Mann= 5 ,-1 , 0
       0     .12       0   396.5    .016       0  418.18     .12       0
   431.1    .045       0   558.6     .12       0
Bank Sta=431.1,558.6
XS Rating Curve= 0 ,0
Exp/Cntr=0.3,0.1

Type RM Length L Ch R = 1 ,47640.3 ,577.1,573.8,570.3
XS GIS Cut Line= 4
     1810858.237      175963.159     1811061.596      176114.579
     1811509.672      176252.953     1811766.441      176240.428
#Sta/Elev= 30
       0 1884.35      39 1872.82    58.5 1867.55      78 1862.99   126.8 1852.86
   204.8 1835.64   273.1 1822.72   302.4 1816.52  318.631813.469   331.7 1811.76
   344.1  1810.7  402.011807.321   419.6 1806.18   439.2 1803.67     576 1803.57
   585.7 1803.74   595.5 1805.29     615 1813.92   624.8 1815.78   644.3 1815.67
   654.1 1816.11   663.9 1817.01     703 1822.62   712.7 1824.39   722.5 1826.78
   779.6 1844.65   798.7 1851.01   903.4  1891.9   960.5 1913.34   979.6  1919.4
#Mann= 6 ,-1 , 0
       0     .12       0  318.63     .06       0   344.1     .12       0
  402.01    .016       0   439.2    .045       0   585.7     .12       0
Bank Sta=439.2,585.7
XS Rating Curve= 0 ,0
Exp/Cntr=0.3,0.1

Type RM Length L Ch R = 1 ,47066.5 ,629.8,606.3,583
XS GIS Cut Line= 4
     1810580.638       176775.32     1810836.061      176666.148
      1811474.95      176801.564     1811726.552      177023.758
#Sta/Elev= 30
       0 1891.61     9.6 1887.93    19.2  1884.9    86.2 1869.17   172.4 1845.71
   201.2 1838.72   220.3 1834.85     249 1830.05   277.8 1825.94  347.01 1817.14
  384.371812.428   433.7 1805.85   453.2 1803.93   472.7 1803.58   599.4 1803.77
   609.2 1805.98   618.9 1810.83   628.7 1814.36   638.4  1815.4   696.9 1814.76
   765.2    1815   843.1 1814.41   862.6 1815.29   891.9 1819.62   969.2 1833.68
   978.8 1836.14  1055.5 1860.23  1141.8 1886.53  1189.8 1899.27  1266.5  1917.6
#Mann= 5 ,-1 , 0
       0     .12       0  347.01    .016       0  384.37     .12       0
   453.2    .045       0   599.4     .12       0
Bank Sta=453.2,599.4
XS Rating Curve= 0 ,0
Exp/Cntr=0.3,0.1

Type RM Length L Ch R = 1 ,46460.2 ,544.2,545.8,547.4
XS GIS Cut Line= 3
     1810770.861      177480.582     1811114.679        177324.8
     1811725.562      177058.153
#Sta/Elev= 30
       0 1925.41    19.4 1918.56    48.4 1906.96    96.8 1889.55   174.2 1860.55
  288.94 1820.63  313.891811.738   329.1 1806.24   338.8 1803.88   348.4 1802.98
   426.5 1801.99  439.241802.872   446.1 1804.02   465.7 1808.94   475.5 1810.31
   544.1 1814.56   563.7 1814.51   661.7 1808.89   681.3  1809.4   700.9 1811.46
   710.7 1813.23   720.5    1816   730.3 1819.58   838.2 1863.02   857.8 1870.32
     946 1898.79  1004.8  1916.9  1024.4    1922  1034.2 1923.63    1044 1924.51
#Mann= 5 ,-1 , 0
       0     .12       0  288.94    .016       0  313.89     .12       0
   338.8    .045       0  439.24     .12       0
Bank Sta=338.8,439.24
XS Rating Curve= 0 ,0
Exp/Cntr=0.3,0.1

Type RM Length L Ch R = 1 ,45914.4 ,498.4,503.5,508.4
XS GIS Cut Line= 2
     1810970.527      177960.336     1811830.745      177625.132
#Sta/Elev= 30
       0 1926.02     9.8 1922.37    29.5  1914.5    68.8 1897.94     108 1882.26
   147.3 1865.62   176.8 1853.97   186.6 1850.52   196.4 1847.63   225.9 1840.84
   245.5 1836.02     275 1827.87   284.8 1825.44  324.221816.975   353.6 1810.67
   363.4 1808.09  372.781805.295     383 1802.51   392.9 1801.44   402.7 1801.38
   530.4 1801.39  539.331801.563     550 1802.32   608.9  1809.5   648.2 1813.66
     658  1815.4   667.9 1818.28   756.3 1849.12   844.6 1876.96   923.2 1902.65
#Mann= 5 ,-1 , 0
       0     .12       0  324.22    .016       0  372.78     .12       0
   392.9    .045       0  539.33     .12       0
Bank Sta=392.9,539.33
XS Rating Curve= 0 ,0
Exp/Cntr=0.3,0.1

Type RM Length L Ch R = 1 ,45410.9 ,407.2,406.7,406
XS GIS Cut Line= 3
     1811089.886      178382.691     1811559.393       178269.02
     1811998.813      178162.634
#Sta/Elev= 30
       0 1924.27    38.6 1901.94    48.3 1896.75      58 1892.19    77.3 1884.81
    96.6 1878.82   135.3 1867.88   164.2 1858.94   212.6  1842.8   251.2 1829.01
   270.5 1822.76   289.8    1818   323.71811.857   338.2 1809.68   347.8  1809.1
  357.561809.515   376.8 1810.47   386.5    1809   396.1 1805.43   405.8 1801.14
   415.4 1798.88   434.8 1798.48   463.8 1798.56   532.2 1799.98   551.9  1800.5
   571.5 1802.48   650.2 1813.65   679.6 1819.53   748.4 1837.37   935.2 1887.82
#Mann= 5 ,-1 , 0
       0     .12       0   323.7    .016       0  357.56     .12       0
   415.4    .045       0   532.2     .12       0
Bank Sta=415.4,532.2
XS Rating Curve= 0 ,0
Exp/Cntr=0.3,0.1

Type RM Length L Ch R = 1 ,45004.2 ,518.6,528.7,538.8
XS GIS Cut Line= 2
     1811097.845      178808.164      1812119.48      178543.404
#Sta/Elev= 30
       0 1953.07     9.8 1948.36    29.3 1938.32    78.2 1910.64      88 1905.72
    97.7 1901.77   107.5 1898.62   224.8 1863.59   263.8  1850.8   302.9 1839.19
   371.3 1820.53   381.1 1818.23   411.7 1813.15  451.641807.015   488.6 1800.77
   498.4 1799.36   508.2 1798.58   527.7 1798.38     645 1798.56   654.7 1799.16
   693.8 1803.26   752.4 1810.02   830.6 1818.32   879.5 1824.29   928.4 1835.93
   996.8  1851.3  1006.5 1853.02  1016.3 1854.33  1045.6    1857  1055.4 1858.54
#Mann= 5 ,-1 , 0
       0     .12       0   411.7    .016       0  451.64     .12       0
   508.2    .045       0     645     .12       0
Bank Sta=508.2,645
XS Rating Curve= 0 ,0
Exp/Cntr=0.3,0.1

Type RM Length L Ch R = 1 ,44475.6 ,593.4,589.4,585.4
XS GIS Cut Line= 3
     1811086.061       178919.62     1811634.672      179176.564
     1812164.312      179184.059
#Sta/Elev= 30
       0 1951.73    78.2 1913.76    97.7 1905.07   107.5  1901.4   263.8 1846.13
   332.2 1827.75   351.8    1822   361.5 1820.39   371.3 1819.79   410.4 1818.82
   517.9 1820.78   566.7 1820.26   615.6 1817.19   625.4 1816.06  636.681813.802
   654.8  1808.1   674.5  1800.4   684.3 1798.62   694.1 1798.38     802 1798.38
   821.6 1798.96   831.4 1800.76   870.6 1810.43  886.021813.149   939.3 1824.52
   949.1 1827.92   978.6 1839.92  1066.8 1872.72  1086.4 1879.01  1135.5  1893.3
#Mann= 5 ,-1 , 0
       0     .12       0  636.68    .016       0   684.3    .045       0
   821.6     .06       0  886.02     .12       0
Bank Sta=684.3,821.6
XS Rating Curve= 0 ,0
Exp/Cntr=0.3,0.1

Type RM Length L Ch R = 1 ,43886.2 ,621.4,609.7,597
XS GIS Cut Line= 3
     1811063.369      180062.637     1811294.394      179808.509
     1812074.774      179741.285
#Sta/Elev= 30
       0 1916.65    19.6 1910.07   117.8 1881.25  244.421841.936  285.841830.471
   343.4 1816.34   392.4  1808.2   421.8 1805.68  501.381802.094  539.33    1801
   578.4 1800.79   627.4  1798.5   695.9 1798.75   705.7 1800.07   735.1 1807.83
   744.9 1808.53   754.7 1805.98   764.4 1801.79   774.2 1798.92     784 1798.34
   891.7 1798.41   901.5 1799.39   911.3 1804.17   930.9 1820.29  970.331850.443
   979.8 1856.75   989.6 1860.61 1014.051866.325  1107.1 1897.06  1126.7 1904.67
#Mann= 9 ,-1 , 0
       0     .12       0  244.42    .016       0  285.84     .12       0
  501.38    .016       0  539.33     .12       0   774.2    .045       0
   901.5     .12       0  970.33    .016       0 1014.05     .12       0
Bank Sta=774.2,901.5
XS Rating Curve= 0 ,0
Exp/Cntr=0.3,0.1

Type RM Length L Ch R = 1 ,43276.5 ,531.9,500.8,470
XS GIS Cut Line= 2
     1811305.051      180526.362     1812071.694      180209.411
#Sta/Elev= 30
       0 1902.81      39  1888.6    68.3 1878.31   136.6 1856.78   185.4 1840.64
  227.451827.202  263.211816.196     283  1810.5   329.41799.642   331.8 1799.12
   341.6 1798.45   351.4 1798.38     449 1798.34   458.7 1798.61   468.5 1800.04
     488 1803.77   497.8 1805.16   507.5 1806.03   595.3 1810.68   624.6 1812.79
   634.4 1814.11   644.1 1816.52   653.9 1819.67  691.351832.539  702.361836.159
   722.2 1842.84   761.3 1858.57   800.3 1873.73   810.1 1877.32   829.6 1883.12
#Mann= 8 ,-1 , 0
       0     .12       0  227.45    .016       0  263.21     .12       0
   329.4     .08       0   331.8    .045       0   458.7     .12       0
  691.35    .016       0  702.36     .12       0
Bank Sta=331.8,458.7
XS Rating Curve= 0 ,0
Exp/Cntr=0.3,0.1

Type RM Length L Ch R = 1 ,42775.6 ,416.5,408.9,401.3
XS GIS Cut Line= 2
     1811878.514      181081.305      1812135.65      180361.327
#Sta/Elev= 30
       0 1900.72    29.4 1890.61      98 1868.64  250.161822.986   284.2 1813.41
     294 1809.93   313.6 1801.54   323.4 1799.48     343 1798.78   411.7 1798.44
   421.5 1798.46   431.3 1799.22   441.1 1801.54   460.7 1808.58   470.5 1811.27
   480.3 1812.38   490.1 1812.45   558.7 1810.05   578.3 1810.44  591.281811.219
   597.9 1811.82   607.7 1813.58   617.5 1815.93   627.3 1819.49  633.391822.436
   666.5 1839.67   686.1 1848.38   725.3 1864.37   744.9 1871.65   764.5 1878.25
#Mann= 6 ,-1 , 0
       0     .12       0  250.16    .016       0   323.4    .045       0
   431.3     .12       0  591.28    .016       0  633.39     .12       0
Bank Sta=323.4,431.3
XS Rating Curve= 0 ,0
Exp/Cntr=0.3,0.1

Type RM Length L Ch R = 1 ,42366.7 ,465.1,495.9,526.6
XS GIS Cut Line= 2
     1812356.894      181197.398      1812460.68      180468.015
#Sta/Elev= 30
       0 1898.02    29.5 1884.65    58.9 1869.01    68.8 1865.94     108    1859
   127.7 1853.67   225.9 1824.54   245.6 1820.58  266.781816.957   304.5 1810.84
   314.3 1808.78   343.8 1800.96   353.6 1799.72   373.3 1798.86   432.2 1796.35
   451.9 1796.04   461.7 1796.76  474.961800.003   491.2 1804.71     501 1806.96
  513.341808.017   550.1 1807.03   559.9 1807.19   579.6 1809.17   599.2 1812.45
   658.2 1827.73   687.6 1835.99   697.4 1839.31   707.3 1843.28   736.7 1855.69
#Mann= 6 ,-1 , 0
       0     .12       0  266.78    .016       0   373.3    .045       0
   461.7     .12       0  474.96    .016       0  513.34     .12       0
#XS Ineff= 2 , 0
                          511.93         1860.55
Permanent Ineff=
       F       F
Bank Sta=373.3,461.7
XS Rating Curve= 0 ,0
Exp/Cntr=0.3,0.1

Type RM Length L Ch R = 1 ,41870.8 ,424.2,448.8,473.5
XS GIS Cut Line= 2
     1812436.755      181287.675     1813208.429      180731.809
#Sta/Elev= 30
       0 1912.05    68.6 1886.97   127.5 1867.82   137.3 1865.69   166.7 1863.64
   176.5 1861.64   186.3 1858.28   205.9 1849.73   225.5 1842.43  305.71 1818.69
  347.591810.796   372.6 1806.83     402 1804.18   441.2 1796.69     451 1795.74
   460.8 1795.59   578.5 1795.72   588.3 1796.68   598.1 1798.84  608.071801.903
   617.7  1804.9   627.5  1807.1  641.081808.241   666.7 1809.92   715.7 1814.36
   735.3  1816.8   745.1 1818.85   784.4 1830.25   833.4  1842.5     951 1873.43
#Mann= 7 ,-1 , 0
       0     .12       0  305.71    .016       0  347.59     .12       0
     451    .045       0   578.5     .12       0  608.07    .016       0
  641.08     .12       0
Bank Sta=451,578.5
XS Rating Curve= 0 ,0
Exp/Cntr=0.3,0.1

Type RM Length L Ch R = 1 ,41422   ,470.6,497.3,523.9
XS GIS Cut Line= 2
     1812450.644      181332.814     1813377.631      181371.709
#Sta/Elev= 30
       0 1927.31    39.1 1909.12   107.4 1885.12   136.7 1873.52   146.5 1870.82
   156.3 1869.03     166 1866.19   175.8 1861.86   185.6 1856.62   205.1 1844.75
   214.9 1839.91   244.2 1829.68  273.371818.111     293 1811.32  305.191808.037
   312.5  1806.5   332.1 1804.47   468.8 1796.37   498.1 1795.59   644.6 1795.58
   664.1 1795.74   673.9 1797.47   683.6 1802.06   703.2 1814.47   712.9 1819.13
   761.8 1832.24  831.481854.235  877.771868.887   908.3 1878.62   927.8 1885.94
#Mann= 7 ,-1 , 0
       0     .12       0  273.37    .016       0  305.19     .12       0
   498.1    .045       0   664.1     .12       0  831.48    .016       0
  877.77     .12       0
Bank Sta=498.1,664.1
XS Rating Curve= 0 ,0
Exp/Cntr=0.3,0.1

Type RM Length L Ch R = 1 ,40924.7 ,431.3,428.8,426.2
XS GIS Cut Line= 2
     1812429.811      181398.786     1813072.619       182000.43
#Sta/Elev= 30
       0 1923.55     9.8 1919.41     137 1870.25   156.5 1861.76   176.1 1851.38
   205.4  1830.9   215.2  1824.6     225 1819.59   234.8 1815.71   244.6 1812.79
   254.4 1810.53  293.99 1803.83   322.8 1798.16  335.571797.342   420.7 1793.56
     450 1792.79   479.4 1792.68   547.8 1792.84   606.5 1795.16   616.3 1797.94
   626.1  1803.4   635.9 1810.22   645.7 1816.23   655.4 1820.89   684.8 1831.26
   714.1  1840.4   733.7 1844.96   753.3 1848.56   831.5 1859.87   880.4 1868.56
#Mann= 5 ,-1 , 0
       0     .12       0  293.99    .016       0  335.57     .12       0
   420.7    .045       0   606.5     .12       0
Bank Sta=420.7,606.5
XS Rating Curve= 0 ,0
Exp/Cntr=0.3,0.1

Type RM Length L Ch R = 1 ,40495.9 ,428.4,423.6,418.9
XS GIS Cut Line= 2
     1812124.255      181666.148     1812852.577      182258.103
#Sta/Elev= 30
       0 1939.37    29.3 1922.44    68.4 1898.64    97.8 1882.08   173.21837.974
  216.18 1811.27   224.9 1806.18   234.6 1801.33   244.4 1798.13   254.2 1796.58
   322.6 1790.65   332.4 1790.22     406 1790.18   449.7 1790.25   459.5 1790.45
   469.3 1791.16     479  1792.7   508.4 1800.13   518.2 1801.47   576.8 1805.98
   684.4 1812.66   723.5 1815.95   762.6 1820.01   782.1 1821.32   791.9 1823.42
   801.7 1826.88   821.2 1834.62   870.1 1852.69   909.2 1866.64   938.5 1877.68
#Mann= 5 ,-1 , 0
       0     .12       0   173.2    .016       0  216.18     .12       0
   322.6    .045       0   469.3     .12       0
Bank Sta=322.6,469.3
XS Rating Curve= 0 ,0
Exp/Cntr=0.3,0.1

Type RM Length L Ch R = 1 ,40072.3 ,373,380.4,387.7
XS GIS Cut Line= 3
     1811887.673      182060.679     1812253.702      182296.052
     1812652.982      182552.808
#Sta/Elev= 30
       0 1906.42      29  1893.7    38.7 1889.18      87 1865.75   125.7 1847.56
   135.4 1843.46   145.1 1839.97  164.191834.202  206.141822.403   270.8 1804.35
   280.4  1802.3   348.1 1791.98   357.8 1790.89   367.5  1790.3   377.2 1790.18
   473.9 1790.19   483.6 1790.29   493.3 1791.01   512.7 1794.59   522.4 1795.86
   570.8 1800.86   648.3 1809.52   677.4 1812.28   687.1 1813.55   696.8 1815.55
   725.8 1823.39   783.9 1837.35   822.7 1847.84   842.1  1852.7   909.9 1868.47
#Mann= 5 ,-1 , 0
       0     .12       0  164.19    .016       0  206.14     .12       0
   348.1    .045       0   493.3     .12       0
Bank Sta=348.1,493.3
XS Rating Curve= 0 ,0
Exp/Cntr=0.3,0.1

Type RM Length L Ch R = 1 ,39691.9 ,444.1,451.7,459.3
XS GIS Cut Line= 2
     1811733.333      182313.688        1812366.      182923.999
#Sta/Elev= 30
       0 1878.39    19.5 1869.62    48.8 1855.14    68.4 1846.55    87.9 1839.41
  120.87 1829.68   146.5 1822.82  162.641819.109   214.9 1808.25   224.6 1806.64
   234.4 1805.73   332.1 1800.85   341.9 1799.34   361.4 1793.62   371.2 1791.39
   380.9 1790.33   390.7 1790.19   468.8 1791.22   488.4 1792.73   595.8 1803.49
   605.6 1804.59   615.3 1806.54   634.9 1814.09   722.8 1851.88   771.6 1871.48
   791.2 1877.75     840 1889.04   859.5 1894.72   869.3 1899.54   879.1 1907.87
#Mann= 5 ,-1 , 0
       0     .12       0  120.87    .016       0  162.64     .12       0
   371.2    .045       0   488.4     .12       0
Bank Sta=371.2,488.4
XS Rating Curve= 0 ,0
Exp/Cntr=0.3,0.1

Type RM Length L Ch R = 1 ,39240.2 ,545.1,559.8,574.5
XS GIS Cut Line= 2
     1811456.792      182520.358     1811933.789      183211.181
#Sta/Elev= 30
       0 1876.77    29.3 1861.86    68.3 1842.67    87.8 1834.59    97.6 1831.07
   117.1 1824.86   136.7 1819.58   156.2 1815.33     205 1807.78   214.8  1806.6
   283.1 1802.52   429.5 1802.59   439.3 1801.39     449 1798.84   468.6 1792.16
   478.3 1789.56   488.1  1788.5   497.8 1788.43   585.7 1788.64   595.5 1791.01
   624.7 1805.42   673.6 1828.54   751.6 1867.43   761.4 1871.64   771.2 1874.66
   800.4 1880.77   810.2 1883.16     820 1886.45   829.7 1890.65   839.5  1895.4
#Mann= 3 ,-1 , 0
       0     .12       0   478.3    .045       0   595.5     .12       0
Bank Sta=478.3,595.5
XS Rating Curve= 0 ,0
Exp/Cntr=0.3,0.1

Type RM Length L Ch R = 1 ,38680.4 ,463.7,439.4,415.1
XS GIS Cut Line= 4
     1811108.769      182712.016     1811218.005       182857.12
     1811294.394      183287.675       1811414.4      183443.683
#Sta/Elev= 30
       0  1904.4    19.1 1894.63    38.2 1884.08    66.9 1867.78      86 1857.63
    95.6 1853.09   114.7 1844.67   124.3 1840.23   181.6 1813.27   191.3 1809.25
   201.1  1806.2   210.8 1804.18   239.9 1799.75   269.1 1795.63   278.8 1793.65
   298.2 1788.23     308  1786.6   317.7 1786.43   473.1 1786.44     512 1786.76
   521.7 1787.24   531.4 1788.66   541.2 1791.12   560.6 1796.72     580 1801.82
   628.8 1812.88     678 1825.49   707.5  1832.7   746.8 1842.79   815.7 1861.49
#Mann= 3 ,-1 , 0
       0     .12       0     308    .045       0     512     .12       0
Bank Sta=308,512
XS Rating Curve= 0 ,0
Exp/Cntr=0.3,0.1

Type RM Length L Ch R = 1 ,38241   ,454.8,430.2,405.8
XS GIS Cut Line= 2
     1810670.336      183065.764     1811253.705      183565.795
#Sta/Elev= 30
       0 1908.37    29.2 1895.04    48.6 1885.51    68.1 1875.51   136.2 1839.21
   175.1  1816.8     214 1793.68   223.7 1788.67   233.4 1785.96   243.2 1785.51
     321 1785.55   330.7  1786.2   340.4  1788.2   359.9 1793.83   369.6 1795.92
   379.3  1797.1  448.98 1801.21   501.81804.209   554.4 1807.32     603 1810.55
   612.7 1811.49   632.2 1814.38   641.9 1816.18   651.6 1818.28   661.4 1820.83
   671.1 1823.72     710 1836.34   729.4 1841.86   748.9 1846.91   768.3 1852.47
#Mann= 5 ,-1 , 0
       0     .12       0   233.4    .045       0   330.7     .12       0
  448.98     .06       0   501.8     .12       0
Bank Sta=233.4,330.7
XS Rating Curve= 0 ,0
Exp/Cntr=0.3,0.1

Type RM Length L Ch R = 1 ,37810.8 ,389.9,388.2,386.2
XS GIS Cut Line= 3
     1810368.839      183614.872     1810995.783      183652.259
     1811158.375      183732.765
#Sta/Elev= 30
       0 1854.68    39.2 1845.35    78.5 1836.83   127.6 1827.42   176.6 1817.51
   255.2 1803.51   274.8 1799.63   284.6 1797.42   294.4 1794.88     314 1788.94
   323.8 1786.34   333.7 1785.04   343.5 1784.84   372.9 1785.28   402.4 1785.44
   412.2 1786.78     422 1789.32   431.8 1791.72   441.6 1793.07   451.4 1793.79
   510.3 1797.56   656.7 1805.73   666.2 1806.37   675.8 1807.66   685.4 1810.16
   694.9  1813.9     714 1822.82   723.6 1826.96   752.2 1838.23   809.5 1861.54
#Mann= 3 ,-1 , 0
       0     .12       0     314    .045       0     422     .12       0
Bank Sta=314,422
XS Rating Curve= 0 ,0
Exp/Cntr=0.3,0.1

Type RM Length L Ch R = 1 ,37422.7 ,334.9,324.7,314.5
XS GIS Cut Line= 2
     1810346.681      184021.404     1811124.649       184028.79
#Sta/Elev= 30
       0 1858.41    68.1 1838.47    97.2 1829.31  126.851821.234   176.71808.364
   194.5 1804.68   204.2 1803.66   223.7 1802.64   272.3 1801.15   301.5 1798.48
   311.2 1797.02   320.9  1794.7   340.4 1789.07   359.8 1784.39   369.6  1783.1
   379.3 1782.87   476.5 1783.08   486.2 1783.93     496 1786.29   515.4 1792.68
   525.2 1794.53   612.7 1803.51   622.4 1805.48   632.1 1809.08   709.9 1843.33
   729.4 1852.38   748.8 1862.22   758.6 1866.75   768.3 1870.27     778 1872.89
#Mann= 5 ,-1 , 0
       0     .12       0  126.85    .016       0   176.7     .12       0
   369.6    .045       0   476.5     .12       0
Bank Sta=369.6,476.5
XS Rating Curve= 0 ,0
Exp/Cntr=0.3,0.1

Type RM Length L Ch R = 1 ,37098   ,499,479.5,460.3
XS GIS Cut Line= 4
     1810412.424      184525.457     1810641.616       184388.37
     1811023.561      184287.675     1811147.632      184226.353
#Sta/Elev= 30
       0 1874.17    76.3 1849.52    95.4 1842.81   114.5 1835.65     124 1832.47
   143.1 1826.68   162.1 1821.53   181.2 1816.89   200.3 1812.72   238.4  1805.7
   267.1 1801.45   276.7 1800.61     296 1799.64   305.6 1798.61   315.2 1796.68
   324.9  1793.9   353.8 1784.65   363.4 1782.94     373 1782.62   469.4 1783.02
     479 1783.45   488.6 1785.57   507.9 1793.91   517.6 1795.58   633.2  1801.8
   642.8  1802.4   652.4 1803.79   662.1 1806.64   671.3 1810.22   800.5 1861.69
#Mann= 3 ,-1 , 0
       0     .12       0   353.8    .045       0   488.6     .12       0
Bank Sta=353.8,488.6
XS Rating Curve= 0 ,0
Exp/Cntr=0.3,0.1

Type RM Length L Ch R = 1 ,36618.5 ,382.2,366.5,350.1
XS GIS Cut Line= 2
     1810743.733      185003.076     1811268.696      184484.901
#Sta/Elev= 30
       0  1921.2    68.8 1889.89    98.4 1876.13   108.2 1871.11   147.5 1849.71
     177 1834.17   226.2 1808.67     236 1803.69   255.7 1794.07   265.5 1789.47
   275.4 1785.49   285.2 1783.27     295 1782.43   314.7 1781.92   344.2 1781.57
   363.9 1781.53   383.6 1781.58   393.4 1782.11   403.2 1784.04   413.1 1787.36
   422.9 1789.82   432.7 1791.34   442.6 1792.04   550.8 1798.19   599.9 1801.15
   619.6 1802.57   629.4 1803.95   639.3 1806.38   688.4 1820.51   737.6 1835.12
#Mann= 3 ,-1 , 0
       0     .12       0   285.2    .045       0   393.4     .12       0
Bank Sta=285.2,393.4
XS Rating Curve= 0 ,0
Exp/Cntr=0.3,0.1

Type RM Length L Ch R = 1 ,36252.1 ,332.7,332.6,332.6
XS GIS Cut Line= 2
     1811195.202      185253.668     1811450.713      184591.146
#Sta/Elev= 30
       0 1915.52    29.2 1901.96    68.1 1883.46    87.5 1874.54   126.4 1857.55
   155.6 1843.76   175.1 1835.48   262.6 1799.68   282.1 1792.64   301.5 1786.38
   311.3 1784.05     321  1782.4   330.7 1781.56   340.4 1781.33   437.7 1781.07
   447.4  1781.2   457.2 1781.95   466.9 1784.02   486.4 1789.34   496.1 1791.36
   515.5 1794.68   583.6 1804.54   632.3 1810.62     642 1812.62   651.7 1815.14
   661.4 1818.26   671.2 1822.32   690.6  1832.7   700.4 1837.45   710.1  1841.2
#Mann= 3 ,-1 , 0
       0     .12       0   330.7    .045       0   447.4     .12       0
Bank Sta=330.7,447.4
XS Rating Curve= 0 ,0
Exp/Cntr=0.3,0.1

Type RM Length L Ch R = 1 ,35919.4 ,334.3,337.2,342.3
XS GIS Cut Line= 3
     1811501.925       185379.82      1811640.87      185019.314
     1811781.721      184653.861
#Sta/Elev= 30
       0 1904.76     9.7 1899.33    67.6 1865.17    77.3 1859.78    86.9 1854.96
   106.2 1847.49   154.5 1832.42   202.8  1814.1   212.5  1810.8   222.2 1808.13
   260.8  1799.5   309.1 1789.76   357.4 1781.69     367 1780.64   386.4 1779.97
   474.5 1779.58   484.3 1779.69   494.1 1780.78   513.6 1785.54   533.2 1789.67
   552.8 1793.42   611.6 1803.74   631.1 1807.96   650.7 1813.05   680.1  1821.6
   699.7 1827.89   729.1 1838.19   738.8 1840.87   768.2 1847.92     778 1850.72
#Mann= 3 ,-1 , 0
       0     .12       0     367    .045       0   484.3     .12       0
Bank Sta=367,484.3
XS Rating Curve= 0 ,0
Exp/Cntr=0.3,0.1

Type RM Length L Ch R = 1 ,35582.2 ,336.9,350,360.8
XS GIS Cut Line= 3
     1811768.936      185515.696     1811954.224      185127.107
     1812130.084       184810.37
#Sta/Elev= 30
       0 1880.22    29.4 1872.14    68.5 1860.48    88.1 1854.05   146.8  1833.8
   166.3 1827.76   176.1 1825.06   303.3 1791.95   322.9 1787.03   342.4 1782.52
   352.2 1780.66     362 1779.12   371.8    1778   381.6 1777.46     438 1777.23
   489.2 1777.23     499  1777.7   508.8 1779.81   538.2 1789.32     548 1791.72
   557.8 1793.38   606.8 1798.53   626.3  1800.8   636.1  1802.6   645.9 1805.18
   675.3 1814.33   694.9 1820.65   743.8 1838.15   773.2 1848.49   792.8 1855.17
#Mann= 3 ,-1 , 0
       0     .12       0   371.8    .045       0     499     .12       0
Bank Sta=371.8,499
XS Rating Curve= 0 ,0
Exp/Cntr=0.3,0.1

Type RM Length L Ch R = 1 ,35232.2 ,354,350,346
XS GIS Cut Line= 3
     1811930.688      185628.546     1812234.388      185329.573
     1812489.314      185078.614
#Sta/Elev= 30
       0  1880.3    38.7  1867.1    87.2 1851.18   125.9  1838.8     155 1829.83
   193.7  1818.5   329.3 1780.27     339 1777.76  345.58 1776.79   348.7 1776.33
   358.4  1775.8   426.2 1775.69   435.8 1775.71   445.5 1776.03   455.2 1777.04
   484.2 1782.61   513.2 1788.72   522.8 1790.24   551.8 1793.34   600.2 1798.09
   609.9 1798.76   629.2 1799.58   638.9 1800.71   658.2  1803.9   667.9 1806.08
   687.2 1811.06   716.2 1816.86   725.9 1819.02   735.6 1821.48   783.9 1835.25
#Mann= 3 ,-1 , 0
       0     .12       0  345.58    .045       0   455.2     .12       0
Bank Sta=345.58,455.2
XS Rating Curve= 0 ,0
Exp/Cntr=0.3,0.1

Type RM Length L Ch R = 1 ,34882.2 ,360.4,350,340
XS GIS Cut Line= 3
     1812256.286       185850.52      1812478.37       185579.91
      1812718.17      185287.091
#Sta/Elev= 30
       0  1861.6     9.7 1857.82    48.6  1843.7    77.8 1833.55    97.2  1826.5
   116.7 1820.08     175 1802.67   204.2 1794.25   252.8 1781.83   262.6  1778.8
   272.3 1776.18     282 1775.37   291.7 1775.32   398.6 1775.33   408.3 1775.37
     418 1775.76   427.7 1776.99   466.5 1783.49   476.2 1784.53     515 1786.93
   534.5 1788.53   553.9 1791.15   563.6 1792.88   573.3 1794.94     583 1797.42
   612.1 1805.89   621.8 1808.44   660.6 1817.36     680 1823.39   728.6 1841.68
#Mann= 3 ,-1 , 0
       0     .12       0     282    .045       0     418     .12       0
Bank Sta=282,418
XS Rating Curve= 0 ,0
Exp/Cntr=0.3,0.1

Type RM Length L Ch R = 1 ,34532.2 ,364.1,371.2,378
XS GIS Cut Line= 3
     1812627.254      186091.594     1812762.949       185781.29
     1812926.094      185416.944
#Sta/Elev= 30
       0 1844.37    48.4 1829.64    58.1 1826.59    77.4 1819.83    96.8 1814.14
   116.1 1809.65   164.5 1799.28   183.8  1794.8   203.2  1789.6   232.2  1780.8
   241.9 1778.14   251.6  1776.3   261.3 1775.64   338.7 1775.37   387.4 1775.57
   397.1 1776.33   484.7 1786.32   494.5  1787.9   533.4 1795.85   572.4 1801.87
   591.8 1805.46   601.6  1807.7   611.3 1810.56   630.8 1818.24   650.2 1825.08
   679.5 1833.55   708.7 1842.74   718.4 1846.29   728.1 1850.42   737.9 1855.04
#Mann= 3 ,-1 , 0
       0     .12       0   251.6    .045       0   387.4     .12       0
Bank Sta=251.6,387.4
XS Rating Curve= 0 ,0
Exp/Cntr=0.3,0.1

Type RM Length L Ch R = 1 ,34160.9 ,407.2,411.7,416.1
XS GIS Cut Line= 2
     1812852.133      186260.079     1813302.214      185601.942
#Sta/Elev= 30
       0  1834.6    5.121833.122    29.2 1826.53   59.841819.022    87.5 1812.73
    97.2 1811.16   194.5 1799.56   330.6 1784.02   340.3 1782.58     350 1780.51
   369.5 1775.56   379.2 1773.79   388.9 1772.91   408.4 1772.63   515.3 1772.76
   525.1 1773.81   534.8 1776.07   554.2 1781.49   593.1  1791.4     632 1803.39
   651.5 1810.07   661.2 1813.79   670.9 1817.87   680.6 1822.47   690.4 1827.59
   709.8 1838.33   719.5 1842.81   748.7 1854.87   787.6 1870.51   797.3 1874.64
#Mann= 5 ,-1 , 0
       0     .12       0    5.12    .016       0   59.84     .12       0
   388.9    .045       0   515.3     .12       0
Bank Sta=388.9,515.3
XS Rating Curve= 0 ,0
Exp/Cntr=0.3,0.1

Type RM Length L Ch R = 1 ,33749.3 ,523.5,551.1,578.7
XS GIS Cut Line= 4
     1813029.069      186481.651     1813242.311      186343.231
     1813575.644      185961.286     1813658.288      185746.867
#Sta/Elev= 30
       0 1848.98    19.6 1843.84    48.9 1834.19      88 1822.74   127.1 1811.98
     176 1799.49   205.3 1795.84   283.5 1787.65     342 1784.38  376.671783.081
  409.791782.112   527.2 1779.25   566.2 1772.45   585.7 1771.42   644.2 1771.74
   653.9  1772.5   663.7 1774.58   692.9 1783.54   702.7 1784.82   731.9 1784.86
   741.7 1786.86   751.4 1790.96   799.5 1816.62   837.8 1835.43   847.4 1841.02
   885.6 1867.55   943.1 1904.44   952.7 1909.63   962.2 1913.94     991 1925.44
#Mann= 5 ,-1 , 0
       0     .12       0  376.67    .016       0  409.79     .12       0
   566.2    .045       0   653.9     .12       0
#XS Ineff= 2 , 0
                          709.44            1859
Permanent Ineff=
       F       F
Bank Sta=566.2,653.9
XS Rating Curve= 0 ,0
Exp/Cntr=0.3,0.1

Type RM Length L Ch R = 1 ,33198.2 ,362,380.3,398.6
XS GIS Cut Line= 4
     1813129.928      186674.385     1813353.422      186551.564
       1814006.2      186464.759     1814188.368      186543.858
#Sta/Elev= 30
       0 1861.72    19.6  1853.9    39.2 1847.89    88.3  1837.2   137.3 1825.24
   245.2 1796.64   264.8 1793.41   353.3 1781.97  371.391780.628  422.151779.609
  475.431779.036   628.5 1778.64   648.2 1776.63   677.6 1771.28   687.5  1770.9
   766.1 1771.05   775.9 1772.31   785.8 1775.95   815.3  1788.8   834.9 1796.32
   854.6 1801.94   893.9 1811.59   913.5 1817.42   951.4  1830.4   970.3 1834.42
   979.7 1837.36   998.7 1846.18  1008.1 1849.58  1036.5 1858.02  1112.1 1883.59
#Mann= 6 ,-1 , 0
       0     .12       0  371.39     .06       0  422.15    .016       0
  475.43     .12       0   677.6    .045       0   775.9     .12       0
Bank Sta=677.6,775.9
XS Rating Curve= 0 ,0
Exp/Cntr=0.3,0.1

Type RM Length L Ch R = 1 ,32817.8 ,400.4,406.8,413.2
XS GIS Cut Line= 3
     1813165.761       186807.55     1813447.172      186749.481
     1814082.713      186983.628
#Sta/Elev= 30
       0 1879.71    28.7 1870.21   114.9 1840.42   134.1 1833.24   210.7  1803.2
   220.3 1800.05   239.4 1794.73   258.6 1790.37   268.2 1788.98   287.3 1787.45
     356  1784.1   444.4 1781.09   522.9 1779.76   532.7 1779.27   542.6 1777.72
     572  1770.2   581.8  1769.1   591.6 1768.87   660.4 1769.37   670.2 1771.01
     680 1775.72   689.8 1782.19   699.6 1788.13   709.4 1792.67   748.7 1806.95
     788 1818.93   817.4 1826.03   925.4 1850.03     945 1853.54   964.6 1856.45
#Mann= 3 ,-1 , 0
       0     .12       0     572    .045       0   670.2     .12       0
Bank Sta=572,670.2
XS Rating Curve= 0 ,0
Exp/Cntr=0.3,0.1

Type RM Length L Ch R = 1 ,32411   ,393.7,403.9,414.2
XS GIS Cut Line= 2
     1813138.849      186976.178     1813863.036      187393.553
#Sta/Elev= 30
       0 1891.48    19.7 1883.04    98.3 1847.94   196.7 1806.41   226.2 1792.59
   255.7 1777.75   265.5 1773.47   275.3 1770.71   285.2 1770.02     413 1776.18
   432.7  1776.8   442.5 1775.95   452.3 1773.66     472 1768.38   481.8 1766.87
   491.7 1766.43   560.5 1766.27   570.4 1766.49   580.2 1768.19     590 1772.86
   609.7 1785.92   619.5 1790.48   658.8  1803.5   698.2 1814.06   727.7 1822.37
   776.8 1838.22   796.5 1844.26   806.4  1847.7     826 1856.11   835.8 1859.91
#Mann= 3 ,-1 , 0
       0     .12       0     472    .045       0   580.2     .12       0
Bank Sta=472,580.2
XS Rating Curve= 0 ,0
Exp/Cntr=0.3,0.1

Type RM Length L Ch R = 1 ,32007.2 ,398.2,413.1,427.7
XS GIS Cut Line= 2
     1812992.571      187197.472     1813554.638      187776.658
#Sta/Elev= 30
       0 1885.33    98.4 1833.16   118.1 1823.05   147.6 1809.62   216.5 1779.37
   226.4 1775.45   236.2 1772.58   246.1 1771.69   255.9 1771.64   295.3  1772.7
     374 1774.07   383.8 1773.45   393.7 1772.09   413.4 1767.41   423.2 1766.18
   433.1    1766   472.4 1766.07   521.6 1766.71   531.5 1767.74   541.3 1771.21
     561 1782.66   570.9 1787.12   580.7 1789.93   610.2 1795.18   669.3 1805.05
     689 1808.77   698.8 1810.97   738.2 1821.44   777.6  1832.6   807.1 1841.31
#Mann= 3 ,-1 , 0
       0     .12       0   413.4    .045       0   531.5     .12       0
Bank Sta=413.4,531.5
XS Rating Curve= 0 ,0
Exp/Cntr=0.3,0.1

Type RM Length L Ch R = 1 ,31594   ,435.2,453.2,471.1
XS GIS Cut Line= 2
     1812787.355      187349.879     1813084.056      188074.838
#Sta/Elev= 30
       0 1874.78    19.6 1866.99    29.4  1862.6    39.2 1857.69    78.3 1836.28
    88.1 1831.26    97.9 1826.94   127.3 1816.02   176.2 1796.94     186 1793.86
   195.8 1792.04   215.4 1789.93   225.2 1787.06     235 1782.12   254.6 1770.95
   264.4  1766.2   274.2 1763.97   293.4 1763.64   332.9 1764.32   401.4 1764.39
   489.6 1765.22   499.4 1765.36   509.2 1765.97     519 1767.71   528.7 1770.06
   626.7 1794.47   665.8 1804.88     754 1829.11   773.5 1834.55   783.3 1837.53
#Mann= 3 ,-1 , 0
       0     .12       0   264.4    .045       0   509.2     .12       0
Bank Sta=264.4,509.2
XS Rating Curve= 0 ,0
Exp/Cntr=0.3,0.1

Type RM Length L Ch R = 1 ,31140.8 ,393.5,374.9,356.2
XS GIS Cut Line= 4
     1812430.847      187445.745     1812488.839      187662.675
     1812457.589       188013.37     1812518.168      188241.148
#Sta/Elev= 30
       0 1860.98    29.3  1846.7    68.3 1825.44    87.9 1816.77   126.9 1801.11
   136.7 1798.18   146.4 1796.03   156.2 1794.75   234.3 1791.31   244.1 1790.63
   253.9 1788.99   263.7 1785.75     293 1773.46  315.351765.775   322.4 1764.12
   332.1  1763.3   341.9 1763.23     469 1765.16   478.8 1765.85   488.6 1767.34
   527.7  1776.4   566.8 1784.24   576.6 1785.84   615.9  1790.2     665 1799.58
   704.3 1808.23   723.9 1813.15   763.2 1825.07   802.5 1836.09   812.3 1839.43
#Mann= 3 ,-1 , 0
       0     .12       0  315.35    .045       0     469     .12       0
Bank Sta=315.35,469
XS Rating Curve= 0 ,0
Exp/Cntr=0.3,0.1

Type RM Length L Ch R = 1 ,30766   ,337.6,336.6,335.5
XS GIS Cut Line= 3
     1811985.715       187503.68     1812149.003       187885.42
     1812297.038      188268.811
#Sta/Elev= 30
       0 1901.93    38.6 1883.59    67.6 1870.92    86.9 1861.83   164.2 1823.67
   202.8 1804.23   231.7 1790.47   260.7 1776.13     280 1766.28   289.7 1761.74
   299.3 1759.91   318.6 1759.63   386.2 1759.68   395.9 1760.25   405.5 1761.62
   415.2  1763.4   454.3 1771.32   473.9 1774.78   483.7 1776.12   493.5 1776.96
   522.8  1778.7   591.3 1782.11   630.5 1784.33   659.8 1786.29   669.6 1787.48
   679.4 1789.52   689.2 1792.12   718.5 1800.49   777.2 1818.05   826.2 1833.97
#Mann= 3 ,-1 , 0
       0     .12       0   289.7    .045       0   405.5     .12       0
Bank Sta=289.7,405.5
XS Rating Curve= 0 ,0
Exp/Cntr=0.3,0.1

Type RM Length L Ch R = 1 ,30429.4 ,353.3,349.3,345.4
XS GIS Cut Line= 2
     1811658.968      187620.172     1811997.585      188353.178
#Sta/Elev= 30
       0 1926.65    48.6 1900.69    87.6 1881.21   126.5    1861   175.1 1834.84
   204.3 1819.68     214 1814.06   223.8 1807.92   262.7 1781.31   282.1 1768.92
   291.8 1763.83   301.6 1760.63   311.3 1759.57   389.1 1759.63   398.9 1759.72
   408.6 1760.38   418.3 1762.27     428 1765.08   447.5 1769.48   457.2 1771.39
     467 1772.52   554.5 1777.72   661.5 1783.57     681 1784.72   690.7 1785.64
   700.4 1787.23   710.2 1789.29   749.1 1798.26   778.3 1806.08   807.4 1814.85
#Mann= 3 ,-1 , 0
       0     .12       0   301.6    .045       0   408.6     .12       0
Bank Sta=301.6,408.6
XS Rating Curve= 0 ,0
Exp/Cntr=0.3,0.1

Type RM Length L Ch R = 1 ,30080.1 ,468.8,446.9,425
XS GIS Cut Line= 2
     1811330.118      187815.409     1811740.139      188503.747
#Sta/Elev= 30
       0 1917.65    39.1 1904.12    58.6 1896.98    68.4 1893.13    78.2 1888.58
    87.9 1883.16    97.7 1876.53   107.5 1868.84     127 1852.66   166.1 1823.22
   185.6 1807.54   205.2  1793.4   224.7  1775.6   234.5 1767.81   244.3 1761.97
     254 1759.48   263.8 1758.85   273.6 1758.83     342 1758.84   351.8 1758.95
   361.5 1759.61   381.1 1763.94   390.8 1765.56   400.6 1766.53   508.1 1772.52
   664.4 1783.54   674.2 1784.59   693.7 1788.11   781.7 1805.84   801.2 1810.26
#Mann= 3 ,-1 , 0
       0     .12       0     254    .045       0   361.5     .12       0
Bank Sta=254,361.5
XS Rating Curve= 0 ,0
Exp/Cntr=0.3,0.1

Type RM Length L Ch R = 1 ,29633.2 ,349.7,351,355.4
XS GIS Cut Line= 4
     1811025.666      188084.525     1811082.589      188339.759
     1811468.005      188534.203     1811599.254       188707.79
#Sta/Elev= 30
       0 1852.54     9.7  1846.4    19.4  1842.6    48.4 1836.38    67.8 1831.42
   106.5 1818.46   125.9 1812.84   193.7 1797.23   232.4 1790.28   271.3 1782.75
   281.1 1779.97   310.6 1769.83  342.891759.618   349.8 1757.82   359.6 1756.65
   438.1 1755.47   487.2 1755.35     497 1756.03   506.8 1758.32   516.6 1761.81
   526.4 1763.97   595.1 1768.63   604.9 1770.02   634.3 1775.63   683.4 1781.11
   702.6 1783.96   721.6  1788.4     750 1795.92   787.8 1803.89   910.8 1836.76
#Mann= 4 ,-1 , 0
       0     .12       0  342.89     .08       0   359.6    .045       0
     497     .12       0
Bank Sta=359.6,497
XS Rating Curve= 0 ,0
Exp/Cntr=0.3,0.1

Type RM Length L Ch R = 1 ,29282.2 ,347.2,350,349.8
XS GIS Cut Line= 3
     1810698.641      188509.889     1811132.422       188749.24
     1811454.506      188962.455
#Sta/Elev= 30
       0 1793.15      68 1783.67    97.1 1780.51   145.7 1777.13   223.4 1775.17
   262.3 1773.12   330.3 1767.83   427.4 1759.12  455.551755.854  459.361755.426
   466.3 1754.66   495.4 1753.73     563 1754.22   572.7 1754.56   582.3 1755.99
     592 1759.02   601.7 1763.88   630.6 1782.12   649.9 1792.04   669.2 1800.96
   707.9 1817.92   717.5 1821.55   746.5  1828.4   756.2 1831.16   765.8 1834.88
   775.5 1839.38   804.4 1857.27   814.1 1862.78   823.8 1867.45   881.7 1889.69
#Mann= 5 ,-1 , 0
       0     .12       0  455.55     .06       0  459.36     .08       0
   466.3    .045       0   582.3     .12       0
Bank Sta=466.3,582.3
XS Rating Curve= 0 ,0
Exp/Cntr=0.3,0.1

Type RM Length L Ch R = 1 ,28932.2 ,351.8,350,348.2
XS GIS Cut Line= 3
     1810531.093       188773.53     1810939.759      189041.439
     1811261.881      189252.612
#Sta/Elev= 30
       0 1793.93    29.3 1787.29    39.1 1785.92   166.1 1776.64   263.9 1770.12
   322.5 1766.88   371.4  1765.8   381.2  1765.1   390.9 1763.35   400.7 1760.68
   420.2 1754.35     430 1752.63   449.6 1752.23   527.2 1752.37   536.8 1753.65
   546.4 1756.53     585 1770.26   594.6 1773.93   604.2 1778.09   613.8 1782.88
   652.4 1804.19   681.2 1820.61   719.8 1845.12   729.4  1851.6   748.6 1865.45
   767.9 1878.89   787.2 1891.47   796.8  1897.1   806.4    1902   873.8 1933.79
#Mann= 3 ,-1 , 0
       0     .12       0   420.2    .045       0   536.8     .12       0
Bank Sta=420.2,536.8
XS Rating Curve= 0 ,0
Exp/Cntr=0.3,0.1

Type RM Length L Ch R = 1 ,28582.2 ,385,381.3,377.2
XS GIS Cut Line= 3
     1810365.397      189108.629      1810756.59      189339.576
     1811087.386      189534.866
#Sta/Elev= 30
       0 1790.34      29 1783.67    48.3 1780.51    77.3 1777.38     145  1771.5
   183.6 1768.48   212.6 1766.76     261 1764.49   357.6 1760.98   386.6 1758.87
  415.551755.106   425.3 1753.79   444.6 1751.71   511.9 1750.46   521.5 1751.16
  533.231754.201   540.7 1757.22   588.7 1783.27   617.5 1798.12   665.6 1820.26
   675.2 1825.27   694.4 1837.26     704 1842.01   713.6 1845.88   723.2 1849.06
     752 1855.76   780.8 1866.61   790.4 1869.58   828.8 1878.25   838.4 1880.96
#Mann= 4 ,-1 , 0
       0     .12       0  415.55     .08       0   425.3    .045       0
  533.23     .12       0
Bank Sta=425.3,533.23
XS Rating Curve= 0 ,0
Exp/Cntr=0.3,0.1

Type RM Length L Ch R = 1 ,28200.8 ,314.9,324.3,334
XS GIS Cut Line= 2
     1810223.026      189511.595     1810929.711      189834.957
#Sta/Elev= 30
       0 1781.53    68.9 1773.13    88.5 1770.94     118 1768.48   177.1 1764.12
   186.9 1763.76   206.6 1763.74   285.3 1764.34   295.1 1763.91     305 1762.32
   314.8 1759.67   334.5 1753.71   344.3 1751.11   354.2 1749.27     364 1748.59
   442.7 1748.52   452.5 1748.91   462.4 1752.16   472.2 1757.15     482 1760.81
   501.7  1764.6   511.5 1767.04   521.4 1770.16   550.9 1780.84   570.6  1787.4
   580.4 1790.27   609.9 1797.64   629.6 1803.06   649.3 1809.16   777.2 1849.99
#Mann= 3 ,-1 , 0
       0     .12       0   354.2    .045       0   452.5     .12       0
Bank Sta=354.2,452.5
XS Rating Curve= 0 ,0
Exp/Cntr=0.3,0.1

Type RM Length L Ch R = 1 ,27876.6 ,357.1,369.3,381.4
XS GIS Cut Line= 3
     1810120.396      189762.469     1810228.422      189787.675
     1810731.972      190197.262
#Sta/Elev= 30
       0  1786.7     9.2 1783.02    18.5 1780.11    27.7 1778.42    83.2 1773.07
   179.8 1759.53   189.6 1758.51   199.4 1757.96   268.3 1757.43   278.1 1757.24
     288 1756.58   297.8 1754.87   317.5 1749.23  328.711746.904   337.1 1746.21
     347 1746.13   435.5 1746.33   455.1 1747.01     465 1749.78   484.6 1759.54
   504.3 1768.35   514.2 1772.35   563.3  1790.1   592.8 1801.22   632.2 1814.04
     642 1817.87   661.7 1826.87   671.5 1830.97   691.2 1838.49     760 1861.18
#Mann= 3 ,-1 , 0
       0     .12       0  328.71    .045       0   455.1     .12       0
Bank Sta=328.71,455.1
XS Rating Curve= 0 ,0
Exp/Cntr=0.3,0.1

Type RM Length L Ch R = 1 ,27507.3 ,350.7,347.2,343.3
XS GIS Cut Line= 3
     1810000.329      189930.001     1810270.089       190357.12
     1810439.147      190490.416
#Sta/Elev= 30
       0 1798.76     9.7  1796.2    19.4 1793.31    48.6 1784.09    58.3 1781.26
   106.9 1769.28   126.3 1765.08     136 1763.84   145.7    1763   242.9  1755.4
   252.6 1754.05     272 1748.85   281.7 1746.96   291.4 1746.15   301.2 1746.04
   369.2 1746.12   378.9 1746.37   388.6 1747.12   417.7 1750.35   456.6 1754.11
     476 1756.43   495.5 1759.58     515  1763.8   524.8 1766.61   544.3 1773.54
   563.9 1781.07     603  1796.6   671.5 1823.15   700.9 1834.02   720.5 1840.76
#Mann= 3 ,-1 , 0
       0     .12       0   281.7    .045       0   388.6     .12       0
Bank Sta=281.7,388.6
XS Rating Curve= 0 ,0
Exp/Cntr=0.3,0.1

Type RM Length L Ch R = 1 ,27160.1 ,434.3,401.3,368.6
XS GIS Cut Line= 3
     1809720.733      190187.183     1809999.255       190544.62
     1810152.033      190752.953
#Sta/Elev= 30
       0  1799.1    48.2 1788.82    67.5 1785.59    96.4 1781.49   115.7 1777.51
   154.3 1766.31   183.2  1753.6   192.8 1750.64   202.5 1748.31   212.1 1746.12
   221.8 1744.51   231.4 1743.95     241 1743.94   318.2 1743.96   327.8 1744.29
   356.7  1747.4   424.2 1756.43   481.8 1763.56   529.7 1769.06   577.5    1774
   587.1 1776.38   596.7 1780.44   606.2 1785.34   615.8    1791   625.4 1797.78
   634.9 1805.48   644.5 1812.47   654.1 1817.59   663.6 1820.38   711.5 1831.29
#Mann= 3 ,-1 , 0
       0     .12       0   221.8    .045       0   327.8     .12       0
Bank Sta=221.8,327.8
XS Rating Curve= 0 ,0
Exp/Cntr=0.3,0.1

Type RM Length L Ch R = 1 ,26758.8 ,358.5,331.3,304
XS GIS Cut Line= 4
       1809390.2      190580.346     1809488.839      190697.398
     1809950.644      190714.759     1810103.422      190811.981
#Sta/Elev= 30
       0 1790.59   114.8 1770.98   143.5 1765.84   182.6  1757.7   231.7 1746.41
   241.6 1744.83  255.011743.744   290.7 1742.81   310.4 1741.56   320.2 1741.47
     389 1741.72   402.41742.536   546.4 1753.79   575.9 1756.76   615.2 1761.38
   653.3 1765.05   662.9 1766.42   672.4 1768.96   681.9 1773.03   691.4 1778.22
     701 1786.26   710.5 1798.05     720 1810.53   729.6 1819.62   739.1 1825.35
   748.6 1828.96   758.2 1831.75   767.7 1834.16   777.2 1836.31   796.3 1839.55
#Mann= 4 ,-1 , 0
       0     .12       0  255.01     .06       0   290.7    .045       0
   402.4     .12       0
#XS Ineff= 2 , 0
          245.56 1818.25
Permanent Ineff=
       F       F
Bank Sta=290.7,402.4
XS Rating Curve= 0 ,0
Exp/Cntr=0.3,0.1

Type RM Length L Ch R = 1 ,26427.5 ,282,286.6,291.2
XS GIS Cut Line= 3
     1809502.315       191259.51     1809947.172      190895.314
     1810079.116      190839.759
#Sta/Elev= 30
       0 1814.53    58.5 1790.62      78 1784.04  110.371774.571   126.7 1770.52
   136.4 1768.94  171.861766.061  177.631765.519   194.9 1763.87  239.531758.141
  354.741742.328     380 1739.13   399.5 1738.66   477.5 1739.38   487.2 1739.76
     497 1741.01     536 1748.81   565.2 1755.73   584.5 1762.06     594 1766.41
   603.6  1771.7   613.1 1777.92   622.6 1785.29   651.3 1810.54   660.8  1817.5
   670.4 1823.28   679.9  1828.3   689.4 1832.52     699 1835.56   718.1 1838.88
#Mann= 8 ,-1 , 0
       0     .12       0  110.37    .016       0  171.86     .12       0
  177.63    .016       0  239.53     .12       0  354.74     .08       0
     380    .045       0   477.5     .12       0
Bank Sta=380,477.5
XS Rating Curve= 0 ,0
Exp/Cntr=0.3,0.1

Type RM Length L Ch R = 1 ,26140.9 ,369.7,360,350.3
XS GIS Cut Line= 4
     1809758.819      191488.639     1809884.672      191291.148
     1810152.033      191121.009     1810194.666      190998.438
#Sta/Elev= 30
       0 1823.74     9.8 1819.55    19.5 1814.82    29.3 1810.67      39 1807.16
    87.8 1791.63  119.551781.943   136.6 1777.07   146.4 1774.55   161.81771.123
   197.21764.319  225.641758.227     263 1749.74   305.31738.997     311 1737.62
   320.6  1736.2   330.2 1735.85   435.8 1735.81   445.4    1736   455.1 1737.07
   464.7 1739.21   483.9 1744.36   493.5 1746.23   522.3 1750.81   588.2 1760.48
   606.7  1763.5     616 1765.38   625.2 1767.84   643.8  1774.1   680.9 1788.21
#Mann= 8 ,-1 , 0
       0     .12       0  119.55    .016       0   161.8     .12       0
   197.2    .016       0  225.64     .12       0   305.3     .06       0
   320.6    .045       0   445.4     .12       0
Bank Sta=320.6,445.4
XS Rating Curve= 0 ,0
Exp/Cntr=0.3,0.1

Type RM Length L Ch R = 1 ,25780.9 ,283,280.9,278.8
XS GIS Cut Line= 2
     1810019.053      191714.238     1810479.512       191215.83
#Sta/Elev= 30
       0  1860.7    19.7 1852.18    49.2 1838.21   79.971821.745   122.11797.545
   137.7 1788.22   186.8 1757.89   196.7 1752.65   206.5 1749.44   226.2  1745.3
     236 1742.88   255.7 1736.88   265.5 1734.27   275.4 1732.67   285.2 1732.37
   334.4 1732.23   373.7 1732.27   383.5  1732.6  385.391732.913   393.4 1734.24
     413 1739.68   422.9 1741.78   432.7 1743.09   521.2 1749.36   570.4 1752.35
   599.9 1753.81   609.7 1754.67   619.6 1756.23   658.9 1764.19   678.6 1767.51
#Mann= 5 ,-1 , 0
       0     .12       0   79.97    .016       0   122.1     .12       0
   275.4    .045       0  385.39     .12       0
Bank Sta=275.4,385.39
XS Rating Curve= 0 ,0
Exp/Cntr=0.3,0.1

Type RM Length L Ch R = 1 ,25500   ,365,367.5,370.3
XS GIS Cut Line= 2
     1810261.876      191887.314     1810694.283      191364.938
#Sta/Elev= 30
       0 1841.22   40.771826.766      59 1819.82    68.8  1815.8    78.6 1811.49
    98.3 1801.95   127.8 1786.61   186.7 1755.32   196.6 1750.37   235.9 1733.43
   245.7 1730.72   255.5 1730.08   265.4 1730.03     344 1730.06  352.441730.456
   363.6 1731.82   383.3 1736.16   393.1 1738.08   422.6 1742.37   452.1 1746.19
   461.9  1747.2   491.4 1749.39   501.2  1750.3   520.9 1752.47   540.5 1755.17
   550.4 1756.33   579.8 1758.79   619.2 1763.01   648.6 1766.47   678.1 1770.66
#Mann= 4 ,-1 , 0
       0    .016       0   40.77     .12       0   245.7    .045       0
  352.44     .12       0
Bank Sta=245.7,352.44
XS Rating Curve= 0 ,0
Exp/Cntr=0.3,0.1

Type RM Length L Ch R = 1 ,25132.5 ,416.6,432.3,447.5
XS GIS Cut Line= 4
     1810446.267      192063.456     1810645.089       191982.12
     1810864.405      191750.205     1811021.951      191684.693
#Sta/Elev= 30
       0 1805.22    6.871802.605    87.9 1771.39    97.6 1768.14   117.2 1763.16
   136.7  1757.7   146.5 1755.65     166 1752.57   195.3 1748.37   234.2 1743.14
  262.911738.026   272.8 1735.72   292.2 1730.74   301.9 1729.37   311.5 1728.97
   388.9  1729.3   398.6 1729.41   408.3 1729.83   417.9 1730.82   427.6 1732.22
   456.6 1737.11   485.6 1741.03   495.3 1742.74     505 1745.18     534 1753.33
   590.9 1770.45   638.3 1784.38   647.8 1787.52   657.2    1791   704.6 1810.86
#Mann= 5 ,-1 , 0
       0    .016       0    6.87     .12       0  262.91     .06       0
   301.9    .045       0   408.3     .12       0
Bank Sta=301.9,408.3
XS Rating Curve= 0 ,0
Exp/Cntr=0.3,0.1

Type RM Length L Ch R = 1 ,24700.2 ,318.9,318,319.1
XS GIS Cut Line= 3
      1810597.26       192331.41     1810843.005      192287.675
     1811275.223      192105.124
#Sta/Elev= 30
       0 1775.96      48 1760.29    57.6  1757.5    67.2 1755.56      96 1752.95
     144 1746.63     240 1739.72     318 1735.39  335.111733.444   347.4 1730.52
   366.9 1724.19   376.7 1722.54   392.8 1722.13   425.6 1722.17   435.3 1722.69
   445.1 1724.55   474.4 1732.15     494 1738.03   523.3 1749.33   542.8 1758.83
   552.6 1764.58   562.4 1771.26   591.7 1793.93   601.5 1800.87     621  1812.4
   650.4 1826.68   660.2 1830.34   689.5 1838.28   699.2 1841.42   718.8 1849.51
#Mann= 4 ,-1 , 0
       0     .12       0  335.11     .06       0   366.9    .045       0
   445.1     .12       0
Bank Sta=366.9,445.1
XS Rating Curve= 0 ,0
Exp/Cntr=0.3,0.1

Type RM Length L Ch R = 1 ,24382.2 ,346.5,354.7,360.8
XS GIS Cut Line= 3
     1810664.439      192715.596     1811063.207      192535.507
     1811423.293       192395.41
#Sta/Elev= 30
       0 1789.44    19.4 1783.06    48.6 1772.53    58.3 1769.72    87.5 1762.72
   136.1 1749.71   155.6 1745.43   184.7 1740.55   213.9 1736.68   243.1  1734.2
   301.4 1730.82   369.5 1723.49   388.9 1721.59   398.6  1721.1     445 1720.96
   485.8 1720.96   495.5 1721.37  505.991723.307   514.8 1726.06   534.1 1733.19
   563.1 1745.18   572.8 1749.64   611.4 1768.95   650.1 1787.24   659.7 1791.34
   688.7  1801.5     737 1816.03     766 1826.05   804.6 1842.95   823.9 1853.49
#Mann= 3 ,-1 , 0
       0     .12       0   369.5    .045       0  505.99     .12       0
Bank Sta=369.5,505.99
XS Rating Curve= 0 ,0
Exp/Cntr=0.3,0.1
